--- Churchill_Mapping.prj (project) ---

Proj Title=Churchill River Flood Risk Mapping
Current Plan=p35
Default Exp/Contr=0.3,0.1
SI Units
Geom File=g33
Geom File=g14
Geom File=g15
Geom File=g16
Geom File=g17
Geom File=g18
Geom File=g19
Geom File=g06
Unsteady File=u13
Unsteady File=u14
Unsteady File=u15
Unsteady File=u16
Unsteady File=u17
Unsteady File=u01
Unsteady File=u02
Unsteady File=u03
Unsteady File=u07
Unsteady File=u08
Unsteady File=u09
Unsteady File=u10
Unsteady File=u18
Unsteady File=u19
Unsteady File=u20
Unsteady File=u21
Unsteady File=u22
Unsteady File=u23
Plan File=p31
Plan File=p33
Plan File=p34
Plan File=p35
Plan File=p03
Plan File=p04
Plan File=p05
Plan File=p06
Plan File=p11
Plan File=p12
Plan File=p13
Plan File=p14
Plan File=p19
Plan File=p20
Plan File=p21
Plan File=p22
Plan File=p23
Plan File=p24
Plan File=p25
Plan File=p26
Plan File=p27
Plan File=p28
Plan File=p29
Plan File=p30
Y Axis Title=Elevation
X Axis Title(PF)=Main Channel Distance
X Axis Title(XS)=Station
BEGIN DESCRIPTION:
END DESCRIPTION:
DSS Start Date=01JUL2019
DSS Start Time=00:00
DSS End Date=02JUL2019
DSS End Time=00:00
DSS File=dss
DSS Export Rating Curves= 0
DSS Export Rating Curve Sorted= 0
DSS Export Volume Flow Curves= 0
DXF Filename=ChurchillRiver.
DXF OffsetX= 0
DXF OffsetY= 0
DXF ScaleX= 1
DXF ScaleY= 10

--- Churchill_Mapping.p35 (plan) ---

Plan Title=2019 Clipped
Program Version=4.10
Short Identifier=2019 Clipped
Simulation Date=20May2019,00:00,19Jul2019,00:00
Geom File=g33
Flow File=u16
Subcritical Flow
K Sum by GR= 0
Std Step Tol= 0.003
Critical Tol= 0.003
Num of Std Step Trials= 20
Max Error Tol= 0.1
Flow Tol Ratio= 0.001
Split Flow NTrial= 30
Split Flow Tol= 0.006
Split Flow Ratio= 0.02
Log Output Level= 0
Friction Slope Method= 1
Unsteady Friction Slope Method= 2
Unsteady Bridges Friction Slope Method= 1
Parabolic Critical Depth
Global Vel Dist= 0 , 0 , 0
Global Log Level= 0
CheckData=True
Encroach Param=-1 ,0,0, 0
Computation Interval=1HOUR
Output Interval=1HOUR
Run HTab= 1
Run UNet= 1
Run PostProcess= 1
Run WQNet= 0
UNET Theta= 1
UNET Theta Warmup= 1
UNET ZTol= 0.006
UNET ZSATol= 0.015
UNET MxIter= 20
UNET MaxInSteps= 0
UNET DtIC= 0
UNET DtMin= 0
UNET MaxCRTS= 20
UNET WFStab= 2
UNET SFStab= 1
UNET WFX= 1
UNET SFX= 1
UNET DSS MLevel= 4
UNET DZMax Abort= 30
UNET Convert EG Bridges= 0
UNET Use Existing IB Tables=-1
UNET Froude Reduction=False
UNET Froude Limit= 1
UNET Froude Power= 10
UNET Time Slicing=0,0, 5
UNET Junction Losses=0
Instantaneous Interval=1HOUR
DSS File=dss
Write IC File= 0
Write IC File at Sim End=0
Echo Input=False
Echo Parameters=False
Echo Output=False
Write Detailed= 0
WQ AD Non Conservative
WQ ULTIMATE=-1
WQ Max Comp Step=1HOUR
WQ Output Interval=15MIN
WQ Output Selected Increments= 0
WQ Output face flow=0
WQ Output face velocity=0
WQ Output face area=0
WQ Output face dispersion=0
WQ Output cell volume=0
WQ Output cell surface area=0
WQ Output cell continuity=0
WQ Output cumulative cell continuity=0
WQ Output face conc=0
WQ Output face dconc_dx=0
WQ Output face courant=0
WQ Output face peclet=0
WQ Output face adv mass=0
WQ Output face disp mass=0
WQ Output cell mass=0
WQ Output cell source sink temp=0
WQ Output cell source sink nsm=0
WQ Output MaxMinRange=-1
WQ Daily Max Min Mean=-1
WQ Daily Range=0
WQ Daily Time=0
WQ Create Restart=0
WQ Fixed Restart=0
WQ System Summary=0
WQ Use Fixed Temperature=0
Sorting and Armoring Iterations= 10
XS Update Threshold= 0.02
Hydraulics Update Threshold= 0.02
Energy Slope Method= 1
Volume Change Method= 0
XS Weighting Method= 0
Number of US Weighted Cross Sections= 1
Number of DS Weighted Cross Sections= 1
Upstream XS Weight=0.25
Main XS Weight=0.5
Downstream XS Weight=0.25
Number of DS XS's Weighted with US Boundary= 1
Upstream Boundary Weight= 1
Weight of XSs Associated with US Boundary= 0
Number of US XS's Weighted with DS Boundary= 1
Downstream Boundary Weight= 0.5
Weight of XSs Associated with DS Boundary= 0.5
Sediment Output Level= 4
Mass or Volume Output= 0
Output Increment Type= 1
Profile and TS Output Increment= 10
XS Output Flag= 0
XS Output Increment= 10
Disregard all LS=0
Disregard all Conn=0
Disregard all Breaches=0
Disregard all Pumps=0

--- Churchill_Mapping.p03 (plan) ---

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Plan Title=2018 Jun-Aug
Short Identifier=2018
Simulation Date=01Jun2018,00:00,31Jul2018,00:00
Geom File=g06
Flow File=u17

--- Churchill_Mapping.p04 (plan) ---

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Plan Title=2019
Short Identifier=2019
Geom File=g06
Flow File=u01

--- Churchill_Mapping.p05 (plan) ---

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Plan Title=2017 Oct-Nov
Short Identifier=2017 Fall
Simulation Date=15Oct2017,00:00,14Nov2017,00:00
Geom File=g06
Flow File=u02

--- Churchill_Mapping.p06 (plan) ---

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Plan Title=2017 Jun - Aug
Short Identifier=2017
Simulation Date=15Jun2017,00:00,14Sep2017,00:00
Geom File=g06
Flow File=u03

--- Churchill_Mapping.p11 (plan) ---

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Plan Title=20 Year CLC
Short Identifier=20 YR CLC
Simulation Date=01JUL2019,00:00,31JUL2019,00:00
Geom File=g06
Flow File=u07
Num of Std Step Trials= 40
Split Flow NTrial= 100
Global Vel Dist= 5 , 25 , 5
Optimized Storage Area=Mud Lake
Optimized Weir=Churchill River ,Main            ,4000
Computation Interval=1MIN
UNET ZSATol= 0.006
UNET Froude Limit= 0.8
UNET Froude Power= 4
Volume Change Method= 1
Upstream XS Weight=0
Main XS Weight=1
Downstream XS Weight=0
Sediment Output Level= 3
Profile and TS Output Increment= 1

--- Churchill_Mapping.p12 (plan) ---

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Plan Title=100 Year CLC
Short Identifier=100 YR CLC
Simulation Date=01JUL2019,00:00,31JUL2019,00:00
Geom File=g06
Flow File=u08
Num of Std Step Trials= 40
Split Flow NTrial= 100
Global Vel Dist= 5 , 25 , 5
Optimized Storage Area=Mud Lake
Optimized Weir=Churchill River ,Main            ,4000
Computation Interval=1MIN
UNET ZSATol= 0.006
UNET Froude Limit= 0.8
UNET Froude Power= 4
Volume Change Method= 1
Upstream XS Weight=0
Main XS Weight=1
Downstream XS Weight=0
Sediment Output Level= 3
Profile and TS Output Increment= 1

--- Churchill_Mapping.p13 (plan) ---

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Plan Title=100 Year CC
Short Identifier=100 YR CC
Simulation Date=01JUL2019,00:00,31JUL2019,00:00
Geom File=g06
Flow File=u09
Num of Std Step Trials= 40
Split Flow NTrial= 100
Global Vel Dist= 5 , 25 , 5
Optimized Storage Area=Mud Lake
Optimized Weir=Churchill River ,Main            ,4000
Computation Interval=1MIN
UNET ZSATol= 0.006
UNET Froude Limit= 0.8
UNET Froude Power= 4
Volume Change Method= 1
Upstream XS Weight=0
Main XS Weight=1
Downstream XS Weight=0
Sediment Output Level= 3
Profile and TS Output Increment= 1

--- Churchill_Mapping.p14 (plan) ---

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Plan Title=20 Year CC
Short Identifier=20 YR CC
Simulation Date=01JUL2019,00:00,31JUL2019,00:00
Geom File=g06
Flow File=u10
Num of Std Step Trials= 40
Split Flow NTrial= 100
Global Vel Dist= 5 , 25 , 5
Optimized Storage Area=Mud Lake
Optimized Weir=Churchill River ,Main            ,4000
Computation Interval=1MIN
UNET ZSATol= 0.006
UNET Froude Limit= 0.8
UNET Froude Power= 4
Volume Change Method= 1
Upstream XS Weight=0
Main XS Weight=1
Downstream XS Weight=0
Sediment Output Level= 3
Profile and TS Output Increment= 1

--- Churchill_Mapping.p19 (plan) ---

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Plan Title=Sensitivity_n-30%
Short Identifier=n-30%
Simulation Date=01JUL2019,00:00,02JUL2019,00:00
Geom File=g16
Flow File=u09
Num of Std Step Trials= 40
Split Flow NTrial= 20
Global Vel Dist= 5 , 25 , 5
Optimized Storage Area=Mud Lake
Optimized Weir=Churchill River ,Main            ,4000
Computation Interval=1MIN
Run HTab=-1
Run UNet=-1
Run PostProcess=-1
UNET ZSATol= 0.006
UNET Froude Limit= 0.8
UNET Froude Power= 4
Volume Change Method= 1
Upstream XS Weight=0
Main XS Weight=1
Downstream XS Weight=0
Sediment Output Level= 3
Profile and TS Output Increment= 1

--- Churchill_Mapping.p20 (plan) ---

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Plan Title=Sensitivity_n-20%
Short Identifier=n-20%
Simulation Date=01JUL2019,00:00,31JUL2019,00:00
Geom File=g15
Flow File=u09
Num of Std Step Trials= 40
Split Flow NTrial= 20
Global Vel Dist= 5 , 25 , 5
Optimized Storage Area=Mud Lake
Optimized Weir=Churchill River ,Main            ,4000
Computation Interval=1MIN
Run HTab=-1
Run UNet=-1
Run PostProcess=-1
UNET ZSATol= 0.006
UNET Froude Limit= 0.8
UNET Froude Power= 4
Volume Change Method= 1
Upstream XS Weight=0
Main XS Weight=1
Downstream XS Weight=0
Sediment Output Level= 3
Profile and TS Output Increment= 1

--- Churchill_Mapping.p21 (plan) ---

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Plan Title=Sensitivity_n-10%
Short Identifier=n-10%
Simulation Date=01JUL2019,00:00,31JUL2019,00:00
Geom File=g14
Flow File=u09
Num of Std Step Trials= 40
Split Flow NTrial= 20
Global Vel Dist= 5 , 25 , 5
Optimized Storage Area=Mud Lake
Optimized Weir=Churchill River ,Main            ,4000
Computation Interval=1MIN
Run HTab=-1
Run UNet=-1
Run PostProcess=-1
UNET ZSATol= 0.006
UNET Froude Limit= 0.8
UNET Froude Power= 4
Volume Change Method= 1
Upstream XS Weight=0
Main XS Weight=1
Downstream XS Weight=0
Sediment Output Level= 3
Profile and TS Output Increment= 1

--- Churchill_Mapping.u16 (unsteady flow) ---

Flow Title=2019 Clipped
Program Version=4.10
Use Restart= 0
Initial Flow Loc=Churchill River ,Main            ,41243.44,4321.8
Initial Flow Loc=Churchill River ,Main DS         ,874.7763,4336.9
Initial Flow Loc=Mud Lake A      ,Main A          ,4343.607,7.55
Initial Flow Loc=Mud Lake B      ,Main            ,5538.203,7.55
Initial Flow Loc=Mud Lake C      ,Main            ,3296.746,7.55
Initial Flow Loc=Mud Lake C      ,Main            ,2548.565,15.1
Initial Flow Loc=Mud Lake In     ,In              ,100     ,15.1
Initial Storage Elev=Mud Lake        ,0.5
Boundary Location=Churchill River ,Main            ,41243.44,        ,                ,                ,
Interval=1HOUR
Flow Hydrograph= 1464
  4321.8  4330.6    4326  4327.8    4329  4327.6  4324.3  4302.3  4312.7  4317.5
  4315.8  4316.6  4316.3  4311.8  4310.7  4309.4  4309.6    4310  4304.5  4301.4
  4190.8  4198.4  4197.7  4198.1  4201.4  4199.5  4204.3  4200.4  4201.5  4202.5
  4202.6  4203.7  4201.7  4202.6  4204.7  4202.6  4204.5  4200.8  4193.9  4194.2
  4194.1    4195  4198.9    4197  4192.7  4193.8  4198.3  4199.3  4197.7  4200.4
  4198.6  4202.8  4198.4    4202  4200.2  4201.7  4197.4  4197.3    4197  4193.5
  4191.8  4194.1  4190.3  4109.9    4114  4111.5  4114.5  4113.7    4118  4119.4
    4116  4119.2  4121.9  4123.2  4123.8  4125.6  4125.2  4126.6  4126.7  4130.8
  4129.1  4131.2  4131.4  4132.5  4134.6  4133.7  4132.8  4134.9  4132.8  4131.1
  4131.2  4129.7  4130.7  4128.5  4130.4  4127.3    4131  4132.4  4126.1    4128
    4129  4127.7  4125.6    4124    4127  4120.8  4119.7  4118.3  4118.3  4118.3
  4115.2  4003.9  4003.9  4003.9  4003.9  4003.9  4000.9  4003.9  4003.9  4003.9
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Use DSS=False
CWMS InputPosition= 0
Use Fixed Start Time=False
Is Critical Boundary=False
Boundary Location=Mud Lake In     ,In              ,100     ,        ,                ,                ,
Interval=1HOUR
Flow Hydrograph= 1465
    15.1    15.1    15.2    15.2    15.2    15.3    15.3    15.4    15.4    15.5
    15.5    15.6    15.6    15.6    15.7    15.7    15.8    15.8    15.9    15.9
      16      16      16    16.1    16.1    16.2    16.2    16.3    16.3    16.3
    16.4    16.4    16.5    16.5    16.6    16.6    16.6    16.7    16.7    16.8
    16.8    16.8    16.9    16.9      17      17      17    17.1    17.1    17.2
    17.2    17.2    17.3    17.3    17.4    17.4    17.4    17.5    17.5    17.5
    17.6    17.6    17.6    17.7    17.7    17.8    17.8    17.8    17.9    17.9
    17.9      18      18      18    18.1    18.1    18.1    18.2    18.2    18.2
    18.2    18.3    18.3    18.3    18.4    18.4    18.4    18.5    18.5    18.5
    18.6    18.6    18.6    18.6    18.7    18.7    18.7    18.8    18.8    18.8
    18.8    18.9    18.9    18.9      19      19      19      19    19.1    19.1
    19.1    19.2    19.2    19.2    19.2    19.3    19.3    19.3    19.3    19.4
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Use DSS=False
CWMS InputPosition= 0
Use Fixed Start Time=False
Is Critical Boundary=False
Boundary Location=Churchill River ,Main            ,40242.1 ,        ,                ,                ,
Interval=1HOUR
Lateral Inflow Hydrograph= 1464
    46.7    46.6    46.6    46.5    46.5    46.4    46.3    46.3    46.2    46.2
    46.2    46.1    46.1      46      46      46      46    45.9    45.9    45.9
    45.9    45.9    45.9    45.9    45.8    45.8    45.8    45.8    45.8    45.8
    45.8    45.8    45.8    45.8    45.8    45.8    45.7    45.7    45.7    45.7
    45.6    45.6    45.6    45.5    45.5    45.4    45.4    45.3    45.3    45.2
    45.1      45      45    44.9    44.8    44.8    44.7    44.7    44.6    44.6
    44.6    44.5    44.5    44.5    44.5    44.6    44.6    44.6    44.7    44.7
    44.8    44.9      45    45.1    45.1    45.3    45.4    45.5    45.6    45.7
    45.8      46    46.1    46.2    46.4    46.5    46.6    46.8    46.9      47
    47.2    47.3    47.4    47.5    47.6    47.6    47.7    47.8    47.9      48
      48    48.1    48.2    48.3    48.4    48.5    48.6    48.8    48.9    49.1
    49.3    49.5    49.7      50    50.2    50.5    50.7      51    51.3    51.6
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Use DSS=False
CWMS InputPosition= 0
Use Fixed Start Time=False
Is Critical Boundary=False
Boundary Location=Churchill River ,Main            ,36181.25,        ,                ,                ,
Interval=1HOUR
Lateral Inflow Hydrograph= 1464
    27.2    27.2    27.1    27.1    27.1    27.1    27.1    27.2    27.2    27.3
    27.4    27.5    27.6    27.7    27.8    27.8    27.9    27.9    27.9    27.8
    27.8    27.7    27.6    27.5    27.4    27.3    27.2    27.2    27.1      27
      27      27    26.9    26.9    26.9    26.9    26.8    26.8    26.8    26.8
    26.7    26.6    26.5    26.5    26.4    26.3    26.1      26    25.9    25.8
    25.8    25.7    25.7    25.8    25.9    26.1    26.2    26.5    26.7      27
    27.3    27.6    27.9    28.2    28.3    28.5    28.5    28.5    28.5    28.5
    28.4    28.3    28.3    28.2    28.1      28      28      28      28      28
      28    28.1    28.1    28.2    28.3    28.4    28.5    28.6    28.6    28.5
    28.4    28.3    28.2    28.1    27.9    27.8    27.6    27.5    27.4    27.4
    27.5    27.7      28    28.3    28.7    29.2    29.7    30.3    30.8    31.4
    31.9    32.4    32.7    32.8    32.9    32.9    32.9    32.7    32.5    32.3
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Use DSS=False
CWMS InputPosition= 0
Use Fixed Start Time=False
Is Critical Boundary=False
Boundary Location=Churchill River ,Main            ,25199.9 ,        ,                ,                ,
Interval=1HOUR
Lateral Inflow Hydrograph= 1464
      16      16    15.9    15.9    15.9    15.9      16      16    16.1    16.2
    16.3    16.5    16.6    16.8    16.9    17.1    17.2    17.2    17.3    17.3
    17.3    17.2    17.1    17.1      17    16.9    16.8    16.7    16.6    16.5
    16.5    16.4    16.4    16.4    16.4    16.3    16.3    16.3    16.3    16.3
    16.2    16.1    16.1      16    15.8    15.7    15.6    15.5    15.3    15.2
    15.1    15.1    15.1    15.1    15.2    15.4    15.6    15.9    16.2    16.6
      17    17.4    17.8    18.2    18.5    18.8      19    19.1    19.1    19.1
    19.1    19.1    19.1      19    18.9    18.9    18.9    18.8    18.8    18.9
    18.9      19    19.1    19.2    19.4    19.5    19.7    19.8    19.8    19.8
    19.8    19.7    19.6    19.4    19.3    19.1    18.9    18.7    18.6    18.6
    18.7    18.9    19.2    19.6    20.1    20.7    21.4    22.1    22.9    23.7
    24.4    25.1    25.7    26.1    26.4    26.5    26.6    26.5    26.4    26.2
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Use DSS=False
CWMS InputPosition= 0
Use Fixed Start Time=False
Is Critical Boundary=False
Boundary Location=Churchill River ,Main            ,13613.57,        ,                ,                ,
Interval=1HOUR
Lateral Inflow Hydrograph= 1464
    11.8    11.7    11.7    11.7    11.7    11.7    11.8    11.8    11.9      12
    12.1    12.3    12.4    12.5    12.7    12.7    12.8    12.8    12.8    12.8
    12.8    12.7    12.6    12.5    12.4    12.3    12.2    12.2    12.1    12.1
      12      12      12      12      12      12      12    11.9    11.9    11.9
    11.9    11.8    11.7    11.6    11.5    11.4    11.3    11.2    11.1      11
    10.9    10.9      11      11    11.2    11.4    11.6    11.8    12.1    12.5
    12.9    13.2    13.6    13.9    14.1    14.2    14.3    14.4    14.3    14.3
    14.3    14.2    14.1    14.1      14    13.9    13.9    13.9    13.9    13.9
      14      14    14.1    14.2    14.4    14.5    14.6    14.7    14.7    14.7
    14.6    14.5    14.4    14.2    14.1    13.9    13.7    13.6    13.5    13.5
    13.7    13.9    14.2    14.7    15.1    15.7    16.3    16.9    17.6    18.3
    18.9    19.4    19.7      20    20.1    20.1      20    19.9    19.7    19.4
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Use DSS=False
CWMS InputPosition= 0
Use Fixed Start Time=False
Is Critical Boundary=False
Boundary Location=Churchill River ,Main            ,9566.389,        ,                ,                ,
Interval=1HOUR
Lateral Inflow Hydrograph= 1464
   225.6   225.1   224.6   224.2   223.8   223.4     223   222.7   222.3     222
   221.7   221.5   221.2     221   220.7   220.5   220.4   220.2     220   219.9
   219.7   219.6   219.5   219.3   219.2   219.1     219   218.9   218.8   218.7
   218.6   218.6   218.5   218.4   218.3   218.2   218.1     218     218   217.9
   217.8   217.7   217.5   217.4   217.3   217.2     217   216.8   216.7   216.5
   216.3     216   215.8   215.6   215.4   215.1   214.9   214.7   214.5   214.3
   214.1     214   213.8   213.7   213.6   213.6   213.6   213.6   213.6   213.6
   213.7   213.8   213.9   214.1   214.3   214.5   214.7     215   215.3   215.6
   215.9   216.3   216.7   217.1   217.5     218   218.5     219   219.5     220
   220.5   221.1   221.6   222.2   222.7   223.3   223.8   224.3   224.8   225.3
   225.8   226.3   226.9   227.4   227.9   228.4     229   229.6   230.3     231
   231.7   232.4   233.3   234.1     235   235.9   236.9   237.9   238.9     240
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Use DSS=False
CWMS InputPosition= 0
Use Fixed Start Time=False
Is Critical Boundary=False
Boundary Location=Churchill River ,Main DS         ,32.94778,        ,                ,                ,
Interval=1HOUR
Stage Hydrograph= 1464
    .623    .644    .604    .554    .502    .459    .412    .372    .335    .332
    .337    .383    .451    .468    .469    .427    .382    .341    .304    .271
    .264    .279    .325      .4     .48    .526    .519    .487    .422    .385
     .33     .29    .273    .261    .253    .309    .355    .403    .436    .417
    .381    .337    .308    .274    .249    .251    .265     .32     .39    .469
    .484    .461    .428    .384    .333    .296    .266    .234    .224    .228
    .259    .316    .345    .344    .332    .301    .273    .236    .232    .206
    .202    .228    .262    .332    .392    .407    .381    .342    .303    .283
    .224    .187    .186    .189    .189    .216    .258    .274    .278    .252
    .229    .215    .191    .173    .166    .178    .214    .251    .321     .34
    .345    .327    .303    .268    .234    .216    .205    .193    .198    .213
    .246    .279    .293    .279     .27    .263     .24    .217    .209    .187
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Use DSS=False
CWMS InputPosition= 0
Use Fixed Start Time=False
Is Critical Boundary=False

--- Churchill_Mapping.u01 (unsteady flow) ---

Flow Title=2019
Program Version=4.10
Use Restart= 0
Initial Flow Loc=Churchill River ,Main            ,41243.44,4321.8
Initial Flow Loc=Churchill River ,Main DS         ,874.7763,4336.9
Initial Flow Loc=Mud Lake A      ,Main A          ,4343.607,7.55
Initial Flow Loc=Mud Lake B      ,Main            ,5538.203,7.55
Initial Flow Loc=Mud Lake C      ,Main            ,3296.746,7.55
Initial Flow Loc=Mud Lake C      ,Main            ,2548.565,15.1
Initial Flow Loc=Mud Lake In     ,In              ,100     ,15.1
Initial Storage Elev=Mud Lake        ,0.5
Boundary Location=Churchill River ,Main            ,41243.44,        ,                ,                ,
Interval=1HOUR
Flow Hydrograph= 1464
  4321.8  4330.6    4326  4327.8    4329  4327.6  4324.3  4302.3  4312.7  4317.5
  4315.8  4316.6  4316.3  4311.8  4310.7  4309.4  4309.6    4310  4304.5  4301.4
  4190.8  4198.4  4197.7  4198.1  4201.4  4199.5  4204.3  4200.4  4201.5  4202.5
  4202.6  4203.7  4201.7  4202.6  4204.7  4202.6  4204.5  4200.8  4193.9  4194.2
  4194.1    4195  4198.9    4197  4192.7  4193.8  4198.3  4199.3  4197.7  4200.4
  4198.6  4202.8  4198.4    4202  4200.2  4201.7  4197.4  4197.3    4197  4193.5
  4191.8  4194.1  4190.3  4109.9    4114  4111.5  4114.5  4113.7    4118  4119.4
    4116  4119.2  4121.9  4123.2  4123.8  4125.6  4125.2  4126.6  4126.7  4130.8
  4129.1  4131.2  4131.4  4132.5  4134.6  4133.7  4132.8  4134.9  4132.8  4131.1
  4131.2  4129.7  4130.7  4128.5  4130.4  4127.3    4131  4132.4  4126.1    4128
    4129  4127.7  4125.6    4124    4127  4120.8  4119.7  4118.3  4118.3  4118.3
  4115.2  4003.9  4003.9  4003.9  4003.9  4003.9  4000.9  4003.9  4003.9  4003.9
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Use DSS=False
CWMS InputPosition= 0
Use Fixed Start Time=False
Is Critical Boundary=False
Boundary Location=Mud Lake In     ,In              ,100     ,        ,                ,                ,
Interval=1HOUR
Flow Hydrograph= 1465
    15.1    15.1    15.2    15.2    15.2    15.3    15.3    15.4    15.4    15.5
    15.5    15.6    15.6    15.6    15.7    15.7    15.8    15.8    15.9    15.9
      16      16      16    16.1    16.1    16.2    16.2    16.3    16.3    16.3
    16.4    16.4    16.5    16.5    16.6    16.6    16.6    16.7    16.7    16.8
    16.8    16.8    16.9    16.9      17      17      17    17.1    17.1    17.2
    17.2    17.2    17.3    17.3    17.4    17.4    17.4    17.5    17.5    17.5
    17.6    17.6    17.6    17.7    17.7    17.8    17.8    17.8    17.9    17.9
    17.9      18      18      18    18.1    18.1    18.1    18.2    18.2    18.2
    18.2    18.3    18.3    18.3    18.4    18.4    18.4    18.5    18.5    18.5
    18.6    18.6    18.6    18.6    18.7    18.7    18.7    18.8    18.8    18.8
    18.8    18.9    18.9    18.9      19      19      19      19    19.1    19.1
    19.1    19.2    19.2    19.2    19.2    19.3    19.3    19.3    19.3    19.4
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Use DSS=False
CWMS InputPosition= 0
Use Fixed Start Time=False
Is Critical Boundary=False
Boundary Location=Churchill River ,Main DS         ,-1972.08,        ,                ,                ,
Interval=1HOUR
Stage Hydrograph= 1464
 .163145   .0776   -.024-.137896-.250289 -.35125-.429908-.475389-.476236-.417333
-.318296-.209048-.119516   -.079-.106326-.181488 -.28095-.380572-.456213-.483731
-.442265-.341865-.209249-.071282   .0451.1132438.1100574   .0433   -.065-.193397
-.319491-.421507-.477514-.466956-.395646-.292046-.185242 -.10432   -.077-.106518
-.171999-.252677-.327592-.375779-.376347-.320646-.226243-.114078   -.005   .0797
.1196026.1024795   .0407   -.049 -.15257-.252089-.332164-.376777-.373607-.334506
-.278008-.222355-.185792-.185077-.218146 -.27005-.325589-.369566-.386781-.361677
-.290168-.189693   -.079   .0217   .0946.1202169   .0916   .0225   -.071-.174275
-.270498-.344305-.379971-.368634-.325349-.268073  -.2147-.183124-.188008-.223234
-.274592-.327856-.368804-.383212-.357806-.295912-.212922-.124436   -.046  .00663
   .0185   -.011   -.072-.149825-.232304-.306792-.360592-.381012-.364076-.322722
-.270383-.220492-.186484-.179803-.196312-.225399-.256506-.279075-.282547-.257554
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Use DSS=False
CWMS InputPosition= 0
Use Fixed Start Time=False
Is Critical Boundary=False
Boundary Location=Churchill River ,Main            ,40242.1 ,        ,                ,                ,
Interval=1HOUR
Lateral Inflow Hydrograph= 1464
    46.7    46.6    46.6    46.5    46.5    46.4    46.3    46.3    46.2    46.2
    46.2    46.1    46.1      46      46      46      46    45.9    45.9    45.9
    45.9    45.9    45.9    45.9    45.8    45.8    45.8    45.8    45.8    45.8
    45.8    45.8    45.8    45.8    45.8    45.8    45.7    45.7    45.7    45.7
    45.6    45.6    45.6    45.5    45.5    45.4    45.4    45.3    45.3    45.2
    45.1      45      45    44.9    44.8    44.8    44.7    44.7    44.6    44.6
    44.6    44.5    44.5    44.5    44.5    44.6    44.6    44.6    44.7    44.7
    44.8    44.9      45    45.1    45.1    45.3    45.4    45.5    45.6    45.7
    45.8      46    46.1    46.2    46.4    46.5    46.6    46.8    46.9      47
    47.2    47.3    47.4    47.5    47.6    47.6    47.7    47.8    47.9      48
      48    48.1    48.2    48.3    48.4    48.5    48.6    48.8    48.9    49.1
    49.3    49.5    49.7      50    50.2    50.5    50.7      51    51.3    51.6
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Use DSS=False
CWMS InputPosition= 0
Use Fixed Start Time=False
Is Critical Boundary=False
Boundary Location=Churchill River ,Main            ,36181.25,        ,                ,                ,
Interval=1HOUR
Lateral Inflow Hydrograph= 1464
    27.2    27.2    27.1    27.1    27.1    27.1    27.1    27.2    27.2    27.3
    27.4    27.5    27.6    27.7    27.8    27.8    27.9    27.9    27.9    27.8
    27.8    27.7    27.6    27.5    27.4    27.3    27.2    27.2    27.1      27
      27      27    26.9    26.9    26.9    26.9    26.8    26.8    26.8    26.8
    26.7    26.6    26.5    26.5    26.4    26.3    26.1      26    25.9    25.8
    25.8    25.7    25.7    25.8    25.9    26.1    26.2    26.5    26.7      27
    27.3    27.6    27.9    28.2    28.3    28.5    28.5    28.5    28.5    28.5
    28.4    28.3    28.3    28.2    28.1      28      28      28      28      28
      28    28.1    28.1    28.2    28.3    28.4    28.5    28.6    28.6    28.5
    28.4    28.3    28.2    28.1    27.9    27.8    27.6    27.5    27.4    27.4
    27.5    27.7      28    28.3    28.7    29.2    29.7    30.3    30.8    31.4
    31.9    32.4    32.7    32.8    32.9    32.9    32.9    32.7    32.5    32.3
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Use DSS=False
CWMS InputPosition= 0
Use Fixed Start Time=False
Is Critical Boundary=False
Boundary Location=Churchill River ,Main            ,25199.9 ,        ,                ,                ,
Interval=1HOUR
Lateral Inflow Hydrograph= 1464
      16      16    15.9    15.9    15.9    15.9      16      16    16.1    16.2
    16.3    16.5    16.6    16.8    16.9    17.1    17.2    17.2    17.3    17.3
    17.3    17.2    17.1    17.1      17    16.9    16.8    16.7    16.6    16.5
    16.5    16.4    16.4    16.4    16.4    16.3    16.3    16.3    16.3    16.3
    16.2    16.1    16.1      16    15.8    15.7    15.6    15.5    15.3    15.2
    15.1    15.1    15.1    15.1    15.2    15.4    15.6    15.9    16.2    16.6
      17    17.4    17.8    18.2    18.5    18.8      19    19.1    19.1    19.1
    19.1    19.1    19.1      19    18.9    18.9    18.9    18.8    18.8    18.9
    18.9      19    19.1    19.2    19.4    19.5    19.7    19.8    19.8    19.8
    19.8    19.7    19.6    19.4    19.3    19.1    18.9    18.7    18.6    18.6
    18.7    18.9    19.2    19.6    20.1    20.7    21.4    22.1    22.9    23.7
    24.4    25.1    25.7    26.1    26.4    26.5    26.6    26.5    26.4    26.2
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Use DSS=False
CWMS InputPosition= 0
Use Fixed Start Time=False
Is Critical Boundary=False
Boundary Location=Churchill River ,Main            ,13613.57,        ,                ,                ,
Interval=1HOUR
Lateral Inflow Hydrograph= 1464
    11.8    11.7    11.7    11.7    11.7    11.7    11.8    11.8    11.9      12
    12.1    12.3    12.4    12.5    12.7    12.7    12.8    12.8    12.8    12.8
    12.8    12.7    12.6    12.5    12.4    12.3    12.2    12.2    12.1    12.1
      12      12      12      12      12      12      12    11.9    11.9    11.9
    11.9    11.8    11.7    11.6    11.5    11.4    11.3    11.2    11.1      11
    10.9    10.9      11      11    11.2    11.4    11.6    11.8    12.1    12.5
    12.9    13.2    13.6    13.9    14.1    14.2    14.3    14.4    14.3    14.3
    14.3    14.2    14.1    14.1      14    13.9    13.9    13.9    13.9    13.9
      14      14    14.1    14.2    14.4    14.5    14.6    14.7    14.7    14.7
    14.6    14.5    14.4    14.2    14.1    13.9    13.7    13.6    13.5    13.5
    13.7    13.9    14.2    14.7    15.1    15.7    16.3    16.9    17.6    18.3
    18.9    19.4    19.7      20    20.1    20.1      20    19.9    19.7    19.4
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Use DSS=False
CWMS InputPosition= 0
Use Fixed Start Time=False
Is Critical Boundary=False
Boundary Location=Churchill River ,Main            ,9566.389,        ,                ,                ,
Interval=1HOUR
Lateral Inflow Hydrograph= 1464
   225.6   225.1   224.6   224.2   223.8   223.4     223   222.7   222.3     222
   221.7   221.5   221.2     221   220.7   220.5   220.4   220.2     220   219.9
   219.7   219.6   219.5   219.3   219.2   219.1     219   218.9   218.8   218.7
   218.6   218.6   218.5   218.4   218.3   218.2   218.1     218     218   217.9
   217.8   217.7   217.5   217.4   217.3   217.2     217   216.8   216.7   216.5
   216.3     216   215.8   215.6   215.4   215.1   214.9   214.7   214.5   214.3
   214.1     214   213.8   213.7   213.6   213.6   213.6   213.6   213.6   213.6
   213.7   213.8   213.9   214.1   214.3   214.5   214.7     215   215.3   215.6
   215.9   216.3   216.7   217.1   217.5     218   218.5     219   219.5     220
   220.5   221.1   221.6   222.2   222.7   223.3   223.8   224.3   224.8   225.3
   225.8   226.3   226.9   227.4   227.9   228.4     229   229.6   230.3     231
   231.7   232.4   233.3   234.1     235   235.9   236.9   237.9   238.9     240
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Use DSS=False
CWMS InputPosition= 0
Use Fixed Start Time=False
Is Critical Boundary=False

--- Churchill_Mapping.u02 (unsteady flow) ---

Flow Title=2017 Oct - Nov
Program Version=4.10
Use Restart= 0
Initial Flow Loc=Churchill River ,Main            ,41243.44,1508
Initial Flow Loc=Churchill River ,Main DS         ,874.7763,1511.4
Initial Flow Loc=Mud Lake A      ,Main A          ,4343.607,1.7
Initial Flow Loc=Mud Lake B      ,Main            ,5538.203,1.7
Initial Flow Loc=Mud Lake C      ,Main            ,3296.746,1.7
Initial Flow Loc=Mud Lake C      ,Main            ,2548.565,3.4
Initial Flow Loc=Mud Lake In     ,In              ,100     ,3.4
Initial Storage Elev=Mud Lake        ,0.5
Boundary Location=Churchill River ,Main            ,41243.44,        ,                ,                ,
Interval=1HOUR
Flow Hydrograph= 744
    1508    1507    1507    1507    1507    1508    1507    1507    1507    1507
    1508    1508    1429    1429    1429    1429    1429    1429    1429    1429
    1429    1429    1430    1430    1430    1430    1430    1430    1430    1430
    1430    1431    1431    1431    1431    1431    1432    1432    1432    1432
    1432    1432    1403    1402    1403    1403    1402    1403    1403    1402
    1402    1402    1402    1402    1402    1402    1402    1402    1402    1341
    1341    1341    1342    1342    1342    1341    1342    1342    1341    1341
    1341    1341    1341    1341    1341    1341    1341    1341    1341    1340
    1340    1340    1340    1340    1309    1310    1310    1310    1310    1310
    1310    1311    1311    1311    1311    1311    1311    1311    1311    1312
    1312    1312    1312    1312    1312    1312    1312    1313    1403    1403
    1403    1403    1403    1403    1403    1403    1403    1402    1402    1402
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Use DSS=False
CWMS InputPosition= 0
Use Fixed Start Time=False
Is Critical Boundary=False
Boundary Location=Mud Lake In     ,In              ,100     ,        ,                ,                ,
Interval=1HOUR
Flow Hydrograph= 767
     3.4     3.4     3.4     3.4     3.4     3.4     3.4     3.4     3.4     3.4
     3.4     3.4     3.4     3.4     3.4     3.4     3.4     3.4     3.4     3.4
     3.4     3.4     3.3     3.3     3.3     3.3     3.3     3.3     3.3     3.3
     3.3     3.3     3.3     3.3     3.3     3.3     3.3     3.3     3.3     3.3
     3.3     3.3     3.3     3.3     3.3     3.3     3.3     3.3     3.3     3.3
     3.3     3.3     3.3     3.3     3.3     3.3     3.3     3.3     3.2     3.2
     3.2     3.2     3.2     3.2     3.2     3.2     3.2     3.2     3.2     3.2
     3.2     3.2     3.2     3.2     3.2     3.2     3.2     3.2     3.2     3.2
     3.2     3.2     3.2     3.2     3.2     3.2     3.2     3.2     3.2     3.2
     3.2     3.2     3.2     3.2     3.2     3.1     3.1     3.1     3.1     3.1
     3.1     3.1     3.1     3.1     3.1     3.1     3.1     3.1     3.1     3.1
     3.1     3.1     3.1     3.1     3.1     3.1     3.1     3.1     3.1     3.1
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Use DSS=False
CWMS InputPosition= 0
Use Fixed Start Time=False
Is Critical Boundary=False
Boundary Location=Churchill River ,Main            ,40242.1 ,        ,                ,                ,
Interval=1HOUR
Lateral Inflow Hydrograph= 744
     7.2     7.2     7.3     7.3     7.4     7.4     7.5     7.5     7.6     7.6
     7.7     7.7     7.8     7.8     7.8     7.9     7.9     7.9     7.9       8
       8       8       8       8       8     7.9     7.9     7.9     7.9     7.9
     7.8     7.8     7.8     7.8     7.7     7.7     7.7     7.7     7.6     7.6
     7.6     7.6     7.6     7.6     7.6     7.6     7.6     7.6     7.6     7.6
     7.6     7.6     7.6     7.7     7.7     7.7     7.7     7.7     7.7     7.7
     7.7     7.7     7.7     7.7     7.7     7.7     7.7     7.7     7.7     7.7
     7.7     7.6     7.6     7.6     7.5     7.5     7.5     7.5     7.5     7.5
     7.5     7.5     7.5     7.5     7.4     7.4     7.4     7.4     7.4     7.4
     7.4     7.4     7.4     7.4     7.4     7.4     7.4     7.4     7.4     7.4
     7.3     7.3     7.3     7.3     7.3     7.3     7.3     7.3     7.3     7.3
     7.3     7.3     7.3     7.3     7.3     7.3     7.2     7.2     7.2     7.2
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Use DSS=False
CWMS InputPosition= 0
Use Fixed Start Time=False
Is Critical Boundary=False
Boundary Location=Churchill River ,Main            ,36181.25,        ,                ,                ,
Interval=1HOUR
Lateral Inflow Hydrograph= 744
    23.6    23.6    23.7    23.7    23.7    23.6    23.6    23.5    23.5    23.5
    23.5    23.5    23.4    23.4    23.4    23.4    23.4    23.3    23.3    23.3
    23.3    23.3    23.2    23.2    23.2    23.2    23.2    23.1    23.1    23.1
    23.1    23.1    23.1      23      23      23      23    23.1    23.1    23.2
    23.3    23.4    23.5    23.6    23.6    23.6    23.6    23.6    23.6    23.6
    23.5    23.5    23.5    23.5    23.5    23.4    23.4    23.4    23.4    23.4
    23.3    23.3    23.3    23.3    23.3    23.2    23.2    23.2    23.2    23.2
    23.1    23.1    23.1    23.1    23.1      23      23      23      23      23
    22.9    22.9    22.9    22.9    22.9    22.9    22.8    22.8    22.8    22.8
    22.8    22.8    22.7    22.7    22.7    22.7    22.7    22.7    22.7    22.6
    22.6    22.6    22.6    22.6    22.5    22.5    22.5    22.5    22.5    22.5
    22.4    22.4    22.4    22.4    22.4    22.4    22.3    22.3    22.3    22.3
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Use DSS=False
CWMS InputPosition= 0
Use Fixed Start Time=False
Is Critical Boundary=False
Boundary Location=Churchill River ,Main            ,25199.9 ,        ,                ,                ,
Interval=1HOUR
Lateral Inflow Hydrograph= 744
       7     7.1     7.2     7.2     7.3     7.3     7.2     7.1       7     6.9
     6.8     6.7     6.6     6.5     6.4     6.4     6.3     6.2     6.2     6.2
     6.2     6.2     6.2     6.2     6.2     6.2     6.2     6.2     6.2     6.2
     6.2     6.2     6.2     6.2     6.2     6.2     6.2     6.3     6.3     6.5
     6.6     6.8     6.9       7     7.1     7.2     7.2     7.2     7.1       7
     6.9     6.8     6.7     6.6     6.6     6.5     6.4     6.4     6.3     6.3
     6.2     6.2     6.2     6.2     6.2     6.2     6.2     6.2     6.2     6.2
     6.2     6.2     6.2     6.2     6.2     6.2     6.2     6.2     6.2     6.1
     6.1     6.1     6.1     6.1     6.1     6.1     6.1     6.1     6.1     6.1
     6.1     6.1     6.1     6.1     6.1     6.1     6.1     6.1     6.1     6.1
     6.1     6.1     6.1     6.1     6.1     6.1     6.1     6.1     6.1     6.1
       6       6       6       6       6       6       6       6       6       6
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Use DSS=False
CWMS InputPosition= 0
Use Fixed Start Time=False
Is Critical Boundary=False
Boundary Location=Churchill River ,Main            ,13613.57,        ,                ,                ,
Interval=1HOUR
Lateral Inflow Hydrograph= 744
       5       5     5.1     5.2     5.4     5.6     5.9     6.1     6.4     6.7
       7     7.3     7.6     7.9     8.1     8.3     8.5     8.6     8.6     8.5
     8.3     8.1     7.8     7.5     7.2     6.9     6.6     6.5     6.5     6.5
     6.5     6.5     6.5     6.5     6.5     6.5     6.4     6.4     6.4     6.4
     6.4     6.4     6.4     6.4     6.4     6.4     6.4     6.4     6.4     6.4
     6.4     6.4     6.5     6.5     6.7     6.8     6.9     7.1     7.2     7.3
     7.4     7.5     7.6     7.6     7.7     7.8     7.8     7.8     7.9     7.9
     7.9     7.9     7.9     7.9     7.9     7.9     7.9     7.9     7.9     7.9
     7.9     7.9     7.8     7.7     7.6     7.5     7.4     7.3     7.2       7
     6.9     6.8     6.7     6.6     6.5     6.5     6.5     6.5     6.5     6.5
     6.5     6.5     6.5     6.5     6.4     6.4     6.4     6.4     6.4     6.4
     6.4     6.4     6.4     6.4     6.4     6.4     6.4     6.4     6.4     6.4
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Use DSS=False
CWMS InputPosition= 0
Use Fixed Start Time=False
Is Critical Boundary=False
Boundary Location=Churchill River ,Main            ,9566.389,        ,                ,                ,
Interval=1HOUR
Lateral Inflow Hydrograph= 744
    15.6    15.7    15.8      16    16.1    16.2    16.4    16.5    16.7    16.8
      17    17.2    17.3    17.5    17.6    17.8    17.9    18.1    18.2    18.4
    18.5    18.6    18.7    18.8    18.9      19    19.1    19.2    19.2    19.3
    19.3    19.3    19.4    19.4    19.3    19.3    19.3    19.2    19.2    19.1
    19.1    19.1      19      19      19      19      19    18.9    18.9    18.9
    18.9    18.9    18.8    18.8    18.8    18.8    18.8    18.8    18.8    18.9
    18.9    18.9    18.9    18.9      19      19      19      19      19      19
      19      19    18.9    18.9    18.9    18.8    18.8    18.7    18.7    18.6
    18.6    18.5    18.4    18.3    18.2    18.1      18    17.8    17.7    17.6
    17.5    17.3    17.2    17.1      17    16.9    16.8    16.7    16.6    16.5
    16.4    16.3    16.2    16.1      16      16      16      16    15.9    15.9
    15.9    15.9    15.9    15.9    15.9    15.9    15.8    15.8    15.8    15.8
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Use DSS=False
CWMS InputPosition= 0
Use Fixed Start Time=False
Is Critical Boundary=False
Boundary Location=Churchill River ,Main DS         ,-1972.08,        ,                ,                ,
Interval=1HOUR
Stage Hydrograph= 744
-.216993-.294926-.353979-.380924-.364158-.310257-.237014-.162376-.104291    -.08
-.103121-.159537-.232809-.305787-.361323-.382266-.354053-.284663-.193398   -.099
   -.022   .0178  .00693   -.047-.127895-.218468-.302245-.362552-.382713-.348846
-.271477-.173249   -.076   -.005   .0195-.013127   -.086-.179808-.273557-.347392
-.381173-.357687-.286066-.189374-.090802   -.013   .0192  -.0096   -.087-.193304
-.306294-.405486-.469956-.478779-.420454-.315681-.191924   -.076  .00269   .0208
-.019844   -.098-.195201-.288362-.357493-.381829-.346612 -.26679 -.16641   -.069
 -.00017   .0175   -.027-.116385-.228078-.340495-.431823-.480248-.464672-.385991
-.270578-.146221    -.04   .0181   .0122   -.044-.131296-.228347 -.31522-.371638
 -.37738-.324786-.234671 -.13177    -.04   .0134  .00695    -.06-.164652-.282949
-.391254-.465822-.482914-.422843 -.30232-.154552   -.012   .0897.1204509   .0711
   -.033-.167606-.303891-.415978-.477267-.463207-.380574-.259896-.132223   -.028
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Use DSS=False
CWMS InputPosition= 0
Use Fixed Start Time=False
Is Critical Boundary=False
