HEC-RAS study Churchill_Mapping.prj: Churchill River Flood Risk Mapping

--- Churchill_Mapping.u03 (unsteady flow) ---

Flow Title=2017 Jun - Aug
Program Version=4.10
Use Restart= 0
Initial Flow Loc=Churchill River ,Main            ,41243.44,1458
Initial Flow Loc=Churchill River ,Main DS         ,874.7763,1464.2
Initial Flow Loc=Mud Lake A      ,Main A          ,4343.607,2.6
Initial Flow Loc=Mud Lake B      ,Main            ,5538.203,2.6
Initial Flow Loc=Mud Lake C      ,Main            ,3296.746,2.6
Initial Flow Loc=Mud Lake C      ,Main            ,2548.565,6.2
Initial Flow Loc=Mud Lake In     ,In              ,100     ,6.2
Initial Storage Elev=Mud Lake        ,0.5
Boundary Location=Churchill River ,Main            ,41243.44,        ,                ,                ,
Interval=1HOUR
Flow Hydrograph= 2209
1458.3451459.2141459.2141459.2141459.2141459.2141459.2141459.2141459.2141459.214
1459.2141459.2141459.2141569.3841569.3841569.3841569.3841569.3841569.3841569.384
1569.3841569.3841569.3841569.3841569.3841569.1071569.1071569.1071569.1071569.107
1569.1071569.1071569.1071569.1071569.1071569.1071569.1071588.6281588.6281588.628
1588.6281588.6281588.6281588.6281588.6281588.6281588.6281588.6281588.6281589.781
1589.7811589.7811589.7811589.7811589.7811589.7811589.7811589.7811589.7811589.781
1589.7811589.7811685.0821685.0821685.0821685.0821685.0821685.0821685.0821685.082
1685.0821685.0821685.0821682.4451682.4451682.4451682.4451682.4451682.4451682.445
1682.4451682.4451682.4451682.445 1616.28 1616.28 1616.28 1616.28 1616.28 1616.28
 1616.28 1616.28 1616.28 1616.28 1616.28 1616.28 1616.281617.9541617.9541617.954
1617.9541617.9541617.9541617.9541617.9541617.9541617.9541617.9541617.9541617.954
1617.9541617.9541617.9541617.9541617.9541617.9541617.9541617.9541617.9541617.954
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Use DSS=False
CWMS InputPosition= 0
Use Fixed Start Time=False
Is Critical Boundary=False
Boundary Location=Churchill River ,Main DS         ,32.94778,        ,                ,                ,
Interval=1HOUR
Stage Hydrograph= 2209
   -.023    .075    .152    .173     .16    .119    .056   -.015   -.082   -.147
   -.199   -.227   -.236    -.19    -.13   -.077   -.041   -.055   -.091   -.137
   -.188   -.232    -.25   -.255   -.227   -.168   -.091    -.02    .015    .008
   -.036   -.097    -.16   -.221   -.279   -.317   -.343   -.336   -.283   -.204
   -.151   -.117   -.121   -.155   -.202   -.243   -.269   -.288   -.281   -.246
   -.176   -.109   -.048   -.025   -.034    -.07   -.125   -.185    -.24   -.293
   -.337   -.349   -.337   -.288   -.214   -.145   -.107   -.102   -.142   -.187
   -.222   -.253    -.26   -.265    -.24    -.19   -.107   -.058   -.036   -.048
   -.082   -.124   -.181   -.229   -.267   -.304   -.306   -.281   -.205   -.128
   -.061   -.019   -.012   -.029   -.071   -.111   -.143   -.169   -.175   -.159
   -.109   -.028    .041    .084    .089    .055   -.001   -.048   -.093   -.134
   -.162   -.147   -.105   -.038    .065    .138    .186    .201     .18    .124
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Use DSS=False
CWMS InputPosition= 0
Use Fixed Start Time=False
Is Critical Boundary=False
Boundary Location=Mud Lake In     ,In              ,100     ,        ,                ,                ,
Interval=1HOUR
Flow Hydrograph= 2209
     6.2     6.2     6.2     6.2     6.2     6.2     6.2     6.2     6.2     6.2
     6.2     6.2     6.2     6.2     6.2     6.2     6.2     6.2     6.2     6.2
     6.1     6.1     6.1     6.1     6.1     6.1     6.1     6.1     6.1     6.1
     6.1     6.1     6.1     6.1     6.1     6.1     6.1     6.1     6.1       6
       6       6       6       6       6       6       6       6       6       6
       6       6       6       6       6       6       6       6       6     5.9
     5.9     5.9     5.9     5.9     5.9     5.9     5.9     5.9     5.9     5.9
     5.9     5.9     5.9     5.9     5.9     5.9     5.9     5.9     5.9     5.8
     5.8     5.8     5.8     5.8     5.8     5.8     5.8     5.8     5.8     5.8
     5.8     5.8     5.8     5.8     5.8     5.8     5.8     5.8     5.8     5.8
     5.7     5.7     5.7     5.7     5.7     5.7     5.7     5.7     5.7     5.7
     5.7     5.7     5.7     5.7     5.7     5.7     5.7     5.7     5.7     5.7
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Use DSS=False
CWMS InputPosition= 0
Use Fixed Start Time=False
Is Critical Boundary=False
Boundary Location=Churchill River ,Main            ,40242.1 ,        ,                ,                ,
Interval=1HOUR
Lateral Inflow Hydrograph= 2209
    17.4    17.5    17.6    17.6    17.6    17.6    17.6    17.5    17.4    17.3
    17.1      17    16.8    16.6    16.5    16.3    16.1    15.9    15.7    15.5
    15.4    15.2      15    14.9    14.7    14.6    14.4    14.3    14.2      14
    13.9    13.8    13.7    13.6    13.5    13.4    13.3    13.2    13.1      13
    12.9    12.8    12.7    12.6    12.5    12.4    12.3    12.2    12.1    11.9
    11.8    11.7    11.6    11.5    11.4    11.3    11.2    11.1    10.9    10.8
    10.7    10.6    10.5    10.4    10.3    10.2    10.1      10     9.9     9.8
     9.7     9.6     9.5     9.5     9.4     9.3     9.2     9.1       9       9
     8.9     8.8     8.7     8.7     8.6     8.5     8.5     8.4     8.3     8.3
     8.2     8.2     8.1       8       8     7.9     7.9     7.8     7.8     7.8
     7.8     7.7     7.7     7.7     7.7     7.7     7.7     7.7     7.7     7.7
     7.7     7.7     7.8     7.9       8     8.2     8.4     8.6     8.9     9.2
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Use DSS=False
CWMS InputPosition= 0
Use Fixed Start Time=False
Is Critical Boundary=False
Boundary Location=Churchill River ,Main            ,36181.25,        ,                ,                ,
Interval=1HOUR
Lateral Inflow Hydrograph= 2209
    25.2      25      25      25    24.9    24.9    24.9    24.9    24.9    24.8
    24.8    24.8    24.8    24.7    24.7    24.7    24.7    24.7    24.8    24.8
    24.9      25      25      25    25.1    25.1    25.1    25.1    25.1      25
      25      25    24.9    24.9    24.9    24.9    24.9    24.8    24.8    24.8
    24.8    24.7    24.7    24.7    24.7    24.7    24.6    24.6    24.6    24.6
    24.6    24.5    24.5    24.5    24.5    24.5    24.4    24.4    24.4    24.4
    24.4    24.3    24.3    24.3    24.3    24.3    24.2    24.2    24.2    24.2
    24.2    24.1    24.1    24.1    24.1    24.1      24      24      24      24
    23.9    23.9    23.9    23.9    23.9    23.8    23.8    23.8    23.8    23.8
    23.7    23.7    23.7    23.7    23.7    23.7    23.8    23.9    24.1    24.2
    24.4    24.4    24.5    24.5    24.4    24.4    24.4    24.4    24.4    24.3
    24.5    24.9    25.7    26.7      28    29.4    30.8    31.9    32.8    33.4
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Use DSS=False
CWMS InputPosition= 0
Use Fixed Start Time=False
Is Critical Boundary=False
Boundary Location=Churchill River ,Main            ,25199.9 ,        ,                ,                ,
Interval=1HOUR
Lateral Inflow Hydrograph= 2209
     8.7     8.4     8.1     7.9     7.7     7.5     7.3     7.1       7     6.9
     6.7     6.6     6.5     6.5     6.4     6.4     6.3     6.4     6.4     6.5
     6.6     6.6     6.7     6.8     6.9     6.9     6.9     6.9     6.9     6.9
     6.8     6.7     6.6     6.5     6.4     6.3     6.2     6.2     6.2     6.2
     6.2     6.2     6.2     6.2     6.2     6.2     6.2     6.2     6.2     6.2
     6.2     6.2     6.2     6.2     6.2     6.1     6.1     6.1     6.1     6.1
     6.1     6.1     6.1     6.1     6.1     6.1     6.1     6.1     6.1     6.1
     6.1     6.1     6.1     6.1     6.1       6       6       6       6       6
       6       6       6       6       6       6       6       6       6       6
       6       6       6       6       6       6     6.1     6.3     6.5     6.7
     6.9       7     7.1     7.2     7.2     7.1       7     6.9     6.8     6.8
     6.9     7.4     8.2     9.3    10.8    12.5    14.3      16    17.5    18.6
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Use DSS=False
CWMS InputPosition= 0
Use Fixed Start Time=False
Is Critical Boundary=False
Boundary Location=Churchill River ,Main            ,13613.57,        ,                ,                ,
Interval=1HOUR
Lateral Inflow Hydrograph= 2209
     7.7     7.5     7.3     7.2     7.1     6.9     6.8     6.7     6.7     6.6
     6.5     6.5     6.5     6.5     6.5     6.5     6.5     6.5     6.6     6.7
     6.8     6.9     6.9       7     7.1     7.1     7.1     7.2     7.1     7.1
       7     6.9     6.8     6.7     6.6     6.6     6.5     6.5     6.5     6.5
     6.5     6.5     6.5     6.5     6.5     6.4     6.4     6.4     6.4     6.4
     6.4     6.4     6.4     6.4     6.4     6.4     6.4     6.4     6.4     6.4
     6.4     6.4     6.4     6.4     6.3     6.3     6.3     6.3     6.3     6.3
     6.3     6.3     6.3     6.3     6.3     6.3     6.3     6.3     6.3     6.3
     6.3     6.3     6.3     6.2     6.2     6.2     6.2     6.2     6.2     6.2
     6.2     6.2     6.2     6.2     6.3     6.3     6.4     6.5     6.7     6.9
     7.1     7.2     7.3     7.2     7.2       7     6.9     6.8     6.7     6.7
     6.9     7.5     8.3     9.5      11    12.6    14.2    15.5    16.5    17.2
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Use DSS=False
CWMS InputPosition= 0
Use Fixed Start Time=False
Is Critical Boundary=False
Boundary Location=Churchill River ,Main            ,9566.389,        ,                ,                ,
Interval=1HOUR
Lateral Inflow Hydrograph= 2209
    58.2      59    59.9    60.7    61.4    62.1    62.7    63.2    63.7    64.1
    64.4    64.7    64.9      65    64.9    64.8    64.6    64.3    63.9    63.5
      63    62.5    61.9    61.3    60.6    59.9    59.2    58.5    57.8    57.1
    56.4    55.6    54.9    54.3    53.6    52.9    52.3    51.7    51.1    50.5
    49.9    49.4    48.8    48.3    47.7    47.2    46.7    46.2    45.7    45.2
    44.7    44.2    43.7    43.2    42.7    42.3    41.8    41.3    40.8    40.4
    39.9    39.4      39    38.5      38    37.5      37    36.6    36.1    35.6
    35.2    34.7    34.2    33.8    33.3    32.9    32.5      32    31.6    31.2
    30.8    30.4    30.1    29.7    29.3      29    28.6    28.3    27.9    27.6
    27.3      27    26.6    26.3    26.1    25.8    25.5    25.3      25    24.8
    24.6    24.4    24.2    24.1    23.9    23.8    23.6    23.5    23.4    23.3
    23.2    23.2    23.3    23.5    23.8    24.3    24.8    25.4    26.1      27
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Use DSS=False
CWMS InputPosition= 0
Use Fixed Start Time=False
Is Critical Boundary=False
Boundary Location=Churchill River ,Main DS         ,-1972.08,        ,                ,                ,
Interval=1HOUR
Stage Hydrograph= 2209
-.088874  .00317    .078.1174316.1053915   .0476   -.039-.141688-.241794-.324467
-.373922-.375031-.329945-.257984-.179035-.112983   -.079   -.089-.129984  -.1852
-.239402-.276796-.281586-.241135-.165392   -.072   .0177    .088.1193536   .0986
   .0355   -.054-.156294-.254149-.332753-.376694  -.3721-.324971-.253746-.176916
-.112971    -.08   -.088-.126231-.178548-.231375-.270394-.281288-.253877-.197437
-.126944   -.057  -.0036   .0191.0000269   -.053-.127736-.210583-.288849-.349613
-.379957-.368591-.321178-.253262-.180502-.118553-.083071   -.085-.119371-.169556
-.222642-.264788-.282152-.262334-.209947-.140279   -.068    -.01.0181159  .00403
   -.048-.125883 -.21239-.293668-.355022-.381754-.360687-.297494-.210273-.117327
   -.036   .0125   .0149   -.024    -.09-.164689-.231557-.274179-.276205-.234984
-.167153    -.09   -.023   .0151  .00969   -.039-.116145-.204801-.289226-.353374
-.381204-.359742-.297396-.211638-.119973   -.039.0110633   .0172   -.017   -.078
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Use DSS=False
CWMS InputPosition= 0
Use Fixed Start Time=False
Is Critical Boundary=False

--- Churchill_Mapping.u07 (unsteady flow) ---

Flow Title=20 Year CLC
Program Version=4.10
Use Restart= 0
Initial Flow Loc=Churchill River ,Main            ,41243.44,1508
Initial Flow Loc=Churchill River ,Main DS         ,874.7763,1511.4
Initial Flow Loc=Mud Lake A      ,Main A          ,4343.607,1.7
Initial Flow Loc=Mud Lake B      ,Main            ,5538.203,1.7
Initial Flow Loc=Mud Lake C      ,Main            ,3296.746,3.4
Initial Flow Loc=Mud Lake C      ,Main            ,2548.565,3.4
Initial Flow Loc=Mud Lake In     ,In              ,100     ,3.4
Initial Storage Elev=Mud Lake        ,0.5
Boundary Location=Churchill River ,Main            ,41243.44,        ,                ,                ,
Interval=1HOUR
Flow Hydrograph= 744
  6038.4  6038.4  6038.4  6038.4  6038.4  6038.4  6038.4  6038.4  6038.4  6038.4
  6038.4  6038.4  6038.4  6038.4  6038.4  6038.4  6038.4  6038.4  6038.4  6038.4
  6038.4  6038.4  6038.4  6038.4  6038.4  6038.4  6038.4  6038.4  6038.4  6038.4
  6038.4  6038.4  6038.4  6038.4  6038.4  6038.4  6038.4  6038.4  6038.4  6038.4
  6038.4  6038.4  6038.4  6038.4  6038.4  6038.4  6038.4  6038.4  6038.4  6038.4
  6038.4  6038.4  6038.4  6038.4  6038.4  6038.4  6038.4  6038.4  6038.4  6038.4
  6038.4  6038.4  6038.4  6038.4  6038.4  6038.4  6038.4  6038.4  6038.4  6038.4
  6038.4  6038.4  6038.4  6038.4  6038.4  6038.4  6038.4  6038.4  6038.4  6038.4
  6038.4  6038.4  6038.4  6038.4  6038.4  6038.4  6038.4  6038.4  6038.4  6038.4
  6038.4  6038.4  6038.4  6038.4  6038.4  6038.4  6038.4  6038.4  6038.4  6038.4
  6038.4  6038.4  6038.4  6038.4  6038.4  6038.4  6038.4  6038.4  6038.4  6038.4
  6038.4  6038.4  6038.4  6038.4  6038.4  6038.4  6038.4  6038.4  6038.4  6038.4
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Use DSS=False
CWMS InputPosition= 0
Use Fixed Start Time=False
Is Critical Boundary=False
Boundary Location=Mud Lake In     ,In              ,100     ,        ,                ,                ,
Interval=1HOUR
Flow Hydrograph= 767
   40.49   40.49   40.49   40.49   40.49   40.49   40.49   40.49   40.49   40.49
   40.49   40.49   40.49   40.49   40.49   40.49   40.49   40.49   40.49   40.49
   40.49   40.49   40.49   40.49   40.49   40.49   40.49   40.49   40.49   40.49
   40.49   40.49   40.49   40.49   40.49   40.49   40.49   40.49   40.49   40.49
   40.49   40.49   40.49   40.49   40.49   40.49   40.49   40.49   40.49   40.49
   40.49   40.49   40.49   40.49   40.49   40.49   40.49   40.49   40.49   40.49
   40.49   40.49   40.49   40.49   40.49   40.49   40.49   40.49   40.49   40.49
   40.49   40.49   40.49   40.49   40.49   40.49   40.49   40.49   40.49   40.49
   40.49   40.49   40.49   40.49   40.49   40.49   40.49   40.49   40.49   40.49
   40.49   40.49   40.49   40.49   40.49   40.49   40.49   40.49   40.49   40.49
   40.49   40.49   40.49   40.49   40.49   40.49   40.49   40.49   40.49   40.49
   40.49   40.49   40.49   40.49   40.49   40.49   40.49   40.49   40.49   40.49
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Use DSS=False
CWMS InputPosition= 0
Use Fixed Start Time=False
Is Critical Boundary=False
Boundary Location=Churchill River ,Main            ,40242.1 ,        ,                ,                ,
Interval=1HOUR
Lateral Inflow Hydrograph= 744
   66.98   66.98   66.98   66.98   66.98   66.98   66.98   66.98   66.98   66.98
   66.98   66.98   66.98   66.98   66.98   66.98   66.98   66.98   66.98   66.98
   66.98   66.98   66.98   66.98   66.98   66.98   66.98   66.98   66.98   66.98
   66.98   66.98   66.98   66.98   66.98   66.98   66.98   66.98   66.98   66.98
   66.98   66.98   66.98   66.98   66.98   66.98   66.98   66.98   66.98   66.98
   66.98   66.98   66.98   66.98   66.98   66.98   66.98   66.98   66.98   66.98
   66.98   66.98   66.98   66.98   66.98   66.98   66.98   66.98   66.98   66.98
   66.98   66.98   66.98   66.98   66.98   66.98   66.98   66.98   66.98   66.98
   66.98   66.98   66.98   66.98   66.98   66.98   66.98   66.98   66.98   66.98
   66.98   66.98   66.98   66.98   66.98   66.98   66.98   66.98   66.98   66.98
   66.98   66.98   66.98   66.98   66.98   66.98   66.98   66.98   66.98   66.98
   66.98   66.98   66.98   66.98   66.98   66.98   66.98   66.98   66.98   66.98
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Use DSS=False
CWMS InputPosition= 0
Use Fixed Start Time=False
Is Critical Boundary=False
Boundary Location=Churchill River ,Main            ,36181.25,        ,                ,                ,
Interval=1HOUR
Lateral Inflow Hydrograph= 744
   19.71   19.71   19.71   19.71   19.71   19.71   19.71   19.71   19.71   19.71
   19.71   19.71   19.71   19.71   19.71   19.71   19.71   19.71   19.71   19.71
   19.71   19.71   19.71   19.71   19.71   19.71   19.71   19.71   19.71   19.71
   19.71   19.71   19.71   19.71   19.71   19.71   19.71   19.71   19.71   19.71
   19.71   19.71   19.71   19.71   19.71   19.71   19.71   19.71   19.71   19.71
   19.71   19.71   19.71   19.71   19.71   19.71   19.71   19.71   19.71   19.71
   19.71   19.71   19.71   19.71   19.71   19.71   19.71   19.71   19.71   19.71
   19.71   19.71   19.71   19.71   19.71   19.71   19.71   19.71   19.71   19.71
   19.71   19.71   19.71   19.71   19.71   19.71   19.71   19.71   19.71   19.71
   19.71   19.71   19.71   19.71   19.71   19.71   19.71   19.71   19.71   19.71
   19.71   19.71   19.71   19.71   19.71   19.71   19.71   19.71   19.71   19.71
   19.71   19.71   19.71   19.71   19.71   19.71   19.71   19.71   19.71   19.71
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Use DSS=False
CWMS InputPosition= 0
Use Fixed Start Time=False
Is Critical Boundary=False
Boundary Location=Churchill River ,Main            ,25199.9 ,        ,                ,                ,
Interval=1HOUR
Lateral Inflow Hydrograph= 744
   28.72   28.72   28.72   28.72   28.72   28.72   28.72   28.72   28.72   28.72
   28.72   28.72   28.72   28.72   28.72   28.72   28.72   28.72   28.72   28.72
   28.72   28.72   28.72   28.72   28.72   28.72   28.72   28.72   28.72   28.72
   28.72   28.72   28.72   28.72   28.72   28.72   28.72   28.72   28.72   28.72
   28.72   28.72   28.72   28.72   28.72   28.72   28.72   28.72   28.72   28.72
   28.72   28.72   28.72   28.72   28.72   28.72   28.72   28.72   28.72   28.72
   28.72   28.72   28.72   28.72   28.72   28.72   28.72   28.72   28.72   28.72
   28.72   28.72   28.72   28.72   28.72   28.72   28.72   28.72   28.72   28.72
   28.72   28.72   28.72   28.72   28.72   28.72   28.72   28.72   28.72   28.72
   28.72   28.72   28.72   28.72   28.72   28.72   28.72   28.72   28.72   28.72
   28.72   28.72   28.72   28.72   28.72   28.72   28.72   28.72   28.72   28.72
   28.72   28.72   28.72   28.72   28.72   28.72   28.72   28.72   28.72   28.72
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Use DSS=False
CWMS InputPosition= 0
Use Fixed Start Time=False
Is Critical Boundary=False
Boundary Location=Churchill River ,Main            ,13613.57,        ,                ,                ,
Interval=1HOUR
Lateral Inflow Hydrograph= 744
   22.02   22.02   22.02   22.02   22.02   22.02   22.02   22.02   22.02   22.02
   22.02   22.02   22.02   22.02   22.02   22.02   22.02   22.02   22.02   22.02
   22.02   22.02   22.02   22.02   22.02   22.02   22.02   22.02   22.02   22.02
   22.02   22.02   22.02   22.02   22.02   22.02   22.02   22.02   22.02   22.02
   22.02   22.02   22.02   22.02   22.02   22.02   22.02   22.02   22.02   22.02
   22.02   22.02   22.02   22.02   22.02   22.02   22.02   22.02   22.02   22.02
   22.02   22.02   22.02   22.02   22.02   22.02   22.02   22.02   22.02   22.02
   22.02   22.02   22.02   22.02   22.02   22.02   22.02   22.02   22.02   22.02
   22.02   22.02   22.02   22.02   22.02   22.02   22.02   22.02   22.02   22.02
   22.02   22.02   22.02   22.02   22.02   22.02   22.02   22.02   22.02   22.02
   22.02   22.02   22.02   22.02   22.02   22.02   22.02   22.02   22.02   22.02
   22.02   22.02   22.02   22.02   22.02   22.02   22.02   22.02   22.02   22.02
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Use DSS=False
CWMS InputPosition= 0
Use Fixed Start Time=False
Is Critical Boundary=False
Boundary Location=Churchill River ,Main            ,9566.389,        ,                ,                ,
Interval=1HOUR
Lateral Inflow Hydrograph= 744
  252.37  252.37  252.37  252.37  252.37  252.37  252.37  252.37  252.37  252.37
  252.37  252.37  252.37  252.37  252.37  252.37  252.37  252.37  252.37  252.37
  252.37  252.37  252.37  252.37  252.37  252.37  252.37  252.37  252.37  252.37
  252.37  252.37  252.37  252.37  252.37  252.37  252.37  252.37  252.37  252.37
  252.37  252.37  252.37  252.37  252.37  252.37  252.37  252.37  252.37  252.37
  252.37  252.37  252.37  252.37  252.37  252.37  252.37  252.37  252.37  252.37
  252.37  252.37  252.37  252.37  252.37  252.37  252.37  252.37  252.37  252.37
  252.37  252.37  252.37  252.37  252.37  252.37  252.37  252.37  252.37  252.37
  252.37  252.37  252.37  252.37  252.37  252.37  252.37  252.37  252.37  252.37
  252.37  252.37  252.37  252.37  252.37  252.37  252.37  252.37  252.37  252.37
  252.37  252.37  252.37  252.37  252.37  252.37  252.37  252.37  252.37  252.37
  252.37  252.37  252.37  252.37  252.37  252.37  252.37  252.37  252.37  252.37
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Use DSS=False
CWMS InputPosition= 0
Use Fixed Start Time=False
Is Critical Boundary=False
Boundary Location=Churchill River ,Main DS         ,-1972.08,        ,                ,                ,
Interval=1HOUR
Stage Hydrograph= 744
     .92     .92     .92     .92     .92     .92     .92     .92     .92     .92
     .92     .92     .92     .92     .92     .92     .92     .92     .92     .92
     .92     .92     .92     .92     .92     .92     .92     .92     .92     .92
     .92     .92     .92     .92     .92     .92     .92     .92     .92     .92
     .92     .92     .92     .92     .92     .92     .92     .92     .92     .92
     .92     .92     .92     .92     .92     .92     .92     .92     .92     .92
     .92     .92     .92     .92     .92     .92     .92     .92     .92     .92
     .92     .92     .92     .92     .92     .92     .92     .92     .92     .92
     .92     .92     .92     .92     .92     .92     .92     .92     .92     .92
     .92     .92     .92     .92     .92     .92     .92     .92     .92     .92
     .92     .92     .92     .92     .92     .92     .92     .92     .92     .92
     .92     .92     .92     .92     .92     .92     .92     .92     .92     .92
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Use DSS=False
CWMS InputPosition= 0
Use Fixed Start Time=False
Is Critical Boundary=False

--- Churchill_Mapping.u08 (unsteady flow) ---

Flow Title=100 Year CLC
Program Version=4.10
Use Restart= 0
Initial Flow Loc=Churchill River ,Main            ,41243.44,1508
Initial Flow Loc=Churchill River ,Main DS         ,874.7763,1511.4
Initial Flow Loc=Mud Lake A      ,Main A          ,4343.607,1.7
Initial Flow Loc=Mud Lake B      ,Main            ,5538.203,1.7
Initial Flow Loc=Mud Lake C      ,Main            ,3296.746,3.4
Initial Flow Loc=Mud Lake C      ,Main            ,2548.565,3.4
Initial Flow Loc=Mud Lake In     ,In              ,100     ,3.4
Initial Storage Elev=Mud Lake        ,0.5
Boundary Location=Churchill River ,Main            ,41243.44,        ,                ,                ,
Interval=1HOUR
Flow Hydrograph= 744
  6742.2  6742.2  6742.2  6742.2  6742.2  6742.2  6742.2  6742.2  6742.2  6742.2
  6742.2  6742.2  6742.2  6742.2  6742.2  6742.2  6742.2  6742.2  6742.2  6742.2
  6742.2  6742.2  6742.2  6742.2  6742.2  6742.2  6742.2  6742.2  6742.2  6742.2
  6742.2  6742.2  6742.2  6742.2  6742.2  6742.2  6742.2  6742.2  6742.2  6742.2
  6742.2  6742.2  6742.2  6742.2  6742.2  6742.2  6742.2  6742.2  6742.2  6742.2
  6742.2  6742.2  6742.2  6742.2  6742.2  6742.2  6742.2  6742.2  6742.2  6742.2
  6742.2  6742.2  6742.2  6742.2  6742.2  6742.2  6742.2  6742.2  6742.2  6742.2
  6742.2  6742.2  6742.2  6742.2  6742.2  6742.2  6742.2  6742.2  6742.2  6742.2
  6742.2  6742.2  6742.2  6742.2  6742.2  6742.2  6742.2  6742.2  6742.2  6742.2
  6742.2  6742.2  6742.2  6742.2  6742.2  6742.2  6742.2  6742.2  6742.2  6742.2
  6742.2  6742.2  6742.2  6742.2  6742.2  6742.2  6742.2  6742.2  6742.2  6742.2
  6742.2  6742.2  6742.2  6742.2  6742.2  6742.2  6742.2  6742.2  6742.2  6742.2
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Use DSS=False
CWMS InputPosition= 0
Use Fixed Start Time=False
Is Critical Boundary=False
Boundary Location=Mud Lake In     ,In              ,100     ,        ,                ,                ,
Interval=1HOUR
Flow Hydrograph= 767
    47.8    47.8    47.8    47.8    47.8    47.8    47.8    47.8    47.8    47.8
    47.8    47.8    47.8    47.8    47.8    47.8    47.8    47.8    47.8    47.8
    47.8    47.8    47.8    47.8    47.8    47.8    47.8    47.8    47.8    47.8
    47.8    47.8    47.8    47.8    47.8    47.8    47.8    47.8    47.8    47.8
    47.8    47.8    47.8    47.8    47.8    47.8    47.8    47.8    47.8    47.8
    47.8    47.8    47.8    47.8    47.8    47.8    47.8    47.8    47.8    47.8
    47.8    47.8    47.8    47.8    47.8    47.8    47.8    47.8    47.8    47.8
    47.8    47.8    47.8    47.8    47.8    47.8    47.8    47.8    47.8    47.8
    47.8    47.8    47.8    47.8    47.8    47.8    47.8    47.8    47.8    47.8
    47.8    47.8    47.8    47.8    47.8    47.8    47.8    47.8    47.8    47.8
    47.8    47.8    47.8    47.8    47.8    47.8    47.8    47.8    47.8    47.8
    47.8    47.8    47.8    47.8    47.8    47.8    47.8    47.8    47.8    47.8
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Use DSS=False
CWMS InputPosition= 0
Use Fixed Start Time=False
Is Critical Boundary=False
Boundary Location=Churchill River ,Main            ,40242.1 ,        ,                ,                ,
Interval=1HOUR
Lateral Inflow Hydrograph= 744
78.99471   78.99   78.99   78.99   78.99   78.99   78.99   78.99   78.99   78.99
   78.99   78.99   78.99   78.99   78.99   78.99   78.99   78.99   78.99   78.99
   78.99   78.99   78.99   78.99   78.99   78.99   78.99   78.99   78.99   78.99
   78.99   78.99   78.99   78.99   78.99   78.99   78.99   78.99   78.99   78.99
   78.99   78.99   78.99   78.99   78.99   78.99   78.99   78.99   78.99   78.99
   78.99   78.99   78.99   78.99   78.99   78.99   78.99   78.99   78.99   78.99
   78.99   78.99   78.99   78.99   78.99   78.99   78.99   78.99   78.99   78.99
   78.99   78.99   78.99   78.99   78.99   78.99   78.99   78.99   78.99   78.99
   78.99   78.99   78.99   78.99   78.99   78.99   78.99   78.99   78.99   78.99
   78.99   78.99   78.99   78.99   78.99   78.99   78.99   78.99   78.99   78.99
   78.99   78.99   78.99   78.99   78.99   78.99   78.99   78.99   78.99   78.99
   78.99   78.99   78.99   78.99   78.99   78.99   78.99   78.99   78.99   78.99
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Use DSS=False
CWMS InputPosition= 0
Use Fixed Start Time=False
Is Critical Boundary=False
Boundary Location=Churchill River ,Main            ,36181.25,        ,                ,                ,
Interval=1HOUR
Lateral Inflow Hydrograph= 744
   23.31   23.31   23.31   23.31   23.31   23.31   23.31   23.31   23.31   23.31
   23.31   23.31   23.31   23.31   23.31   23.31   23.31   23.31   23.31   23.31
   23.31   23.31   23.31   23.31   23.31   23.31   23.31   23.31   23.31   23.31
   23.31   23.31   23.31   23.31   23.31   23.31   23.31   23.31   23.31   23.31
   23.31   23.31   23.31   23.31   23.31   23.31   23.31   23.31   23.31   23.31
   23.31   23.31   23.31   23.31   23.31   23.31   23.31   23.31   23.31   23.31
   23.31   23.31   23.31   23.31   23.31   23.31   23.31   23.31   23.31   23.31
   23.31   23.31   23.31   23.31   23.31   23.31   23.31   23.31   23.31   23.31
   23.31   23.31   23.31   23.31   23.31   23.31   23.31   23.31   23.31   23.31
   23.31   23.31   23.31   23.31   23.31   23.31   23.31   23.31   23.31   23.31
   23.31   23.31   23.31   23.31   23.31   23.31   23.31   23.31   23.31   23.31
   23.31   23.31   23.31   23.31   23.31   23.31   23.31   23.31   23.31   23.31
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Use DSS=False
CWMS InputPosition= 0
Use Fixed Start Time=False
Is Critical Boundary=False
Boundary Location=Churchill River ,Main            ,25199.9 ,        ,                ,                ,
Interval=1HOUR
Lateral Inflow Hydrograph= 744
   33.94   33.94   33.94   33.94   33.94   33.94   33.94   33.94   33.94   33.94
   33.94   33.94   33.94   33.94   33.94   33.94   33.94   33.94   33.94   33.94
   33.94   33.94   33.94   33.94   33.94   33.94   33.94   33.94   33.94   33.94
   33.94   33.94   33.94   33.94   33.94   33.94   33.94   33.94   33.94   33.94
   33.94   33.94   33.94   33.94   33.94   33.94   33.94   33.94   33.94   33.94
   33.94   33.94   33.94   33.94   33.94   33.94   33.94   33.94   33.94   33.94
   33.94   33.94   33.94   33.94   33.94   33.94   33.94   33.94   33.94   33.94
   33.94   33.94   33.94   33.94   33.94   33.94   33.94   33.94   33.94   33.94
   33.94   33.94   33.94   33.94   33.94   33.94   33.94   33.94   33.94   33.94
   33.94   33.94   33.94   33.94   33.94   33.94   33.94   33.94   33.94   33.94
   33.94   33.94   33.94   33.94   33.94   33.94   33.94   33.94   33.94   33.94
   33.94   33.94   33.94   33.94   33.94   33.94   33.94   33.94   33.94   33.94
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Use DSS=False
CWMS InputPosition= 0
Use Fixed Start Time=False
Is Critical Boundary=False
Boundary Location=Churchill River ,Main            ,13613.57,        ,                ,                ,
Interval=1HOUR
Lateral Inflow Hydrograph= 744
   26.04   26.04   26.04   26.04   26.04   26.04   26.04   26.04   26.04   26.04
   26.04   26.04   26.04   26.04   26.04   26.04   26.04   26.04   26.04   26.04
   26.04   26.04   26.04   26.04   26.04   26.04   26.04   26.04   26.04   26.04
   26.04   26.04   26.04   26.04   26.04   26.04   26.04   26.04   26.04   26.04
   26.04   26.04   26.04   26.04   26.04   26.04   26.04   26.04   26.04   26.04
   26.04   26.04   26.04   26.04   26.04   26.04   26.04   26.04   26.04   26.04
   26.04   26.04   26.04   26.04   26.04   26.04   26.04   26.04   26.04   26.04
   26.04   26.04   26.04   26.04   26.04   26.04   26.04   26.04   26.04   26.04
   26.04   26.04   26.04   26.04   26.04   26.04   26.04   26.04   26.04   26.04
   26.04   26.04   26.04   26.04   26.04   26.04   26.04   26.04   26.04   26.04
   26.04   26.04   26.04   26.04   26.04   26.04   26.04   26.04   26.04   26.04
   26.04   26.04   26.04   26.04   26.04   26.04   26.04   26.04   26.04   26.04
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Use DSS=False
CWMS InputPosition= 0
Use Fixed Start Time=False
Is Critical Boundary=False
Boundary Location=Churchill River ,Main            ,9566.389,        ,                ,                ,
Interval=1HOUR
Lateral Inflow Hydrograph= 744
  296.69  296.69  296.69  296.69  296.69  296.69  296.69  296.69  296.69  296.69
  296.69  296.69  296.69  296.69  296.69  296.69  296.69  296.69  296.69  296.69
  296.69  296.69  296.69  296.69  296.69  296.69  296.69  296.69  296.69  296.69
  296.69  296.69  296.69  296.69  296.69  296.69  296.69  296.69  296.69  296.69
  296.69  296.69  296.69  296.69  296.69  296.69  296.69  296.69  296.69  296.69
  296.69  296.69  296.69  296.69  296.69  296.69  296.69  296.69  296.69  296.69
  296.69  296.69  296.69  296.69  296.69  296.69  296.69  296.69  296.69  296.69
  296.69  296.69  296.69  296.69  296.69  296.69  296.69  296.69  296.69  296.69
  296.69  296.69  296.69  296.69  296.69  296.69  296.69  296.69  296.69  296.69
  296.69  296.69  296.69  296.69  296.69  296.69  296.69  296.69  296.69  296.69
  296.69  296.69  296.69  296.69  296.69  296.69  296.69  296.69  296.69  296.69
  296.69  296.69  296.69  296.69  296.69  296.69  296.69  296.69  296.69  296.69
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Use DSS=False
CWMS InputPosition= 0
Use Fixed Start Time=False
Is Critical Boundary=False
Boundary Location=Churchill River ,Main DS         ,-1972.08,        ,                ,                ,
Interval=1HOUR
Stage Hydrograph= 744
     .92     .92     .92     .92     .92     .92     .92     .92     .92     .92
     .92     .92     .92     .92     .92     .92     .92     .92     .92     .92
     .92     .92     .92     .92     .92     .92     .92     .92     .92     .92
     .92     .92     .92     .92     .92     .92     .92     .92     .92     .92
     .92     .92     .92     .92     .92     .92     .92     .92     .92     .92
     .92     .92     .92     .92     .92     .92     .92     .92     .92     .92
     .92     .92     .92     .92     .92     .92     .92     .92     .92     .92
     .92     .92     .92     .92     .92     .92     .92     .92     .92     .92
     .92     .92     .92     .92     .92     .92     .92     .92     .92     .92
     .92     .92     .92     .92     .92     .92     .92     .92     .92     .92
     .92     .92     .92     .92     .92     .92     .92     .92     .92     .92
     .92     .92     .92     .92     .92     .92     .92     .92     .92     .92
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Use DSS=False
CWMS InputPosition= 0
Use Fixed Start Time=False
Is Critical Boundary=False

--- Churchill_Mapping.u09 (unsteady flow) ---

Flow Title=100 Year CC
Program Version=4.10
Use Restart= 0
Initial Flow Loc=Churchill River ,Main            ,41243.44,1508
Initial Flow Loc=Churchill River ,Main DS         ,874.7763,1511.4
Initial Flow Loc=Mud Lake A      ,Main A          ,4343.607,1.7
Initial Flow Loc=Mud Lake B      ,Main            ,5538.203,1.7
Initial Flow Loc=Mud Lake C      ,Main            ,3296.746,1.7
Initial Flow Loc=Mud Lake C      ,Main            ,2548.565,3.4
Initial Flow Loc=Mud Lake In     ,In              ,100     ,3.4
Initial Storage Elev=Mud Lake        ,0.5
Boundary Location=Churchill River ,Main            ,41243.44,        ,                ,                ,
Interval=1HOUR
Flow Hydrograph= 744
    6610    6610    6610    6610    6610    6610    6610    6610    6610    6610
    6610    6610    6610    6610    6610    6610    6610    6610    6610    6610
    6610    6610    6610    6610    6610    6610    6610    6610    6610    6610
    6610    6610    6610    6610    6610    6610    6610    6610    6610    6610
    6610    6610    6610    6610    6610    6610    6610    6610    6610    6610
    6610    6610    6610    6610    6610    6610    6610    6610    6610    6610
    6610    6610    6610    6610    6610    6610    6610    6610    6610    6610
    6610    6610    6610    6610    6610    6610    6610    6610    6610    6610
    6610    6610    6610    6610    6610    6610    6610    6610    6610    6610
    6610    6610    6610    6610    6610    6610    6610    6610    6610    6610
    6610    6610    6610    6610    6610    6610    6610    6610    6610    6610
    6610    6610    6610    6610    6610    6610    6610    6610    6610    6610
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Use DSS=False
CWMS InputPosition= 0
Use Fixed Start Time=False
Is Critical Boundary=False
Boundary Location=Mud Lake In     ,In              ,100     ,        ,                ,                ,
Interval=1HOUR
Flow Hydrograph= 767
   46.87   46.87   46.87   46.87   46.87   46.87   46.87   46.87   46.87   46.87
   46.87   46.87   46.87   46.87   46.87   46.87   46.87   46.87   46.87   46.87
   46.87   46.87   46.87   46.87   46.87   46.87   46.87   46.87   46.87   46.87
   46.87   46.87   46.87   46.87   46.87   46.87   46.87   46.87   46.87   46.87
   46.87   46.87   46.87   46.87   46.87   46.87   46.87   46.87   46.87   46.87
   46.87   46.87   46.87   46.87   46.87   46.87   46.87   46.87   46.87   46.87
   46.87   46.87   46.87   46.87   46.87   46.87   46.87   46.87   46.87   46.87
   46.87   46.87   46.87   46.87   46.87   46.87   46.87   46.87   46.87   46.87
   46.87   46.87   46.87   46.87   46.87   46.87   46.87   46.87   46.87   46.87
   46.87   46.87   46.87   46.87   46.87   46.87   46.87   46.87   46.87   46.87
   46.87   46.87   46.87   46.87   46.87   46.87   46.87   46.87   46.87   46.87
   46.87   46.87   46.87   46.87   46.87   46.87   46.87   46.87   46.87   46.87
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Use DSS=False
CWMS InputPosition= 0
Use Fixed Start Time=False
Is Critical Boundary=False
Boundary Location=Churchill River ,Main            ,40242.1 ,        ,                ,                ,
Interval=1HOUR
Lateral Inflow Hydrograph= 744
   77.45   77.45   77.45   77.45   77.45   77.45   77.45   77.45   77.45   77.45
   77.45   77.45   77.45   77.45   77.45   77.45   77.45   77.45   77.45   77.45
   77.45   77.45   77.45   77.45   77.45   77.45   77.45   77.45   77.45   77.45
   77.45   77.45   77.45   77.45   77.45   77.45   77.45   77.45   77.45   77.45
   77.45   77.45   77.45   77.45   77.45   77.45   77.45   77.45   77.45   77.45
   77.45   77.45   77.45   77.45   77.45   77.45   77.45   77.45   77.45   77.45
   77.45   77.45   77.45   77.45   77.45   77.45   77.45   77.45   77.45   77.45
   77.45   77.45   77.45   77.45   77.45   77.45   77.45   77.45   77.45   77.45
   77.45   77.45   77.45   77.45   77.45   77.45   77.45   77.45   77.45   77.45
   77.45   77.45   77.45   77.45   77.45   77.45   77.45   77.45   77.45   77.45
   77.45   77.45   77.45   77.45   77.45   77.45   77.45   77.45   77.45   77.45
   77.45   77.45   77.45   77.45   77.45   77.45   77.45   77.45   77.45   77.45
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Use DSS=False
CWMS InputPosition= 0
Use Fixed Start Time=False
Is Critical Boundary=False
Boundary Location=Churchill River ,Main            ,36181.25,        ,                ,                ,
Interval=1HOUR
Lateral Inflow Hydrograph= 744
   22.85   22.85   22.85   22.85   22.85   22.85   22.85   22.85   22.85   22.85
   22.85   22.85   22.85   22.85   22.85   22.85   22.85   22.85   22.85   22.85
   22.85   22.85   22.85   22.85   22.85   22.85   22.85   22.85   22.85   22.85
   22.85   22.85   22.85   22.85   22.85   22.85   22.85   22.85   22.85   22.85
   22.85   22.85   22.85   22.85   22.85   22.85   22.85   22.85   22.85   22.85
   22.85   22.85   22.85   22.85   22.85   22.85   22.85   22.85   22.85   22.85
   22.85   22.85   22.85   22.85   22.85   22.85   22.85   22.85   22.85   22.85
   22.85   22.85   22.85   22.85   22.85   22.85   22.85   22.85   22.85   22.85
   22.85   22.85   22.85   22.85   22.85   22.85   22.85   22.85   22.85   22.85
   22.85   22.85   22.85   22.85   22.85   22.85   22.85   22.85   22.85   22.85
   22.85   22.85   22.85   22.85   22.85   22.85   22.85   22.85   22.85   22.85
   22.85   22.85   22.85   22.85   22.85   22.85   22.85   22.85   22.85   22.85
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Use DSS=False
CWMS InputPosition= 0
Use Fixed Start Time=False
Is Critical Boundary=False
Boundary Location=Churchill River ,Main            ,25199.9 ,        ,                ,                ,
Interval=1HOUR
Lateral Inflow Hydrograph= 744
   33.27   33.27   33.27   33.27   33.27   33.27   33.27   33.27   33.27   33.27
   33.27   33.27   33.27   33.27   33.27   33.27   33.27   33.27   33.27   33.27
   33.27   33.27   33.27   33.27   33.27   33.27   33.27   33.27   33.27   33.27
   33.27   33.27   33.27   33.27   33.27   33.27   33.27   33.27   33.27   33.27
   33.27   33.27   33.27   33.27   33.27   33.27   33.27   33.27   33.27   33.27
   33.27   33.27   33.27   33.27   33.27   33.27   33.27   33.27   33.27   33.27
   33.27   33.27   33.27   33.27   33.27   33.27   33.27   33.27   33.27   33.27
   33.27   33.27   33.27   33.27   33.27   33.27   33.27   33.27   33.27   33.27
   33.27   33.27   33.27   33.27   33.27   33.27   33.27   33.27   33.27   33.27
   33.27   33.27   33.27   33.27   33.27   33.27   33.27   33.27   33.27   33.27
   33.27   33.27   33.27   33.27   33.27   33.27   33.27   33.27   33.27   33.27
   33.27   33.27   33.27   33.27   33.27   33.27   33.27   33.27   33.27   33.27
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Use DSS=False
CWMS InputPosition= 0
Use Fixed Start Time=False
Is Critical Boundary=False
Boundary Location=Churchill River ,Main            ,13613.57,        ,                ,                ,
Interval=1HOUR
Lateral Inflow Hydrograph= 744
   25.52   25.52   25.52   25.52   25.52   25.52   25.52   25.52   25.52   25.52
   25.52   25.52   25.52   25.52   25.52   25.52   25.52   25.52   25.52   25.52
   25.52   25.52   25.52   25.52   25.52   25.52   25.52   25.52   25.52   25.52
   25.52   25.52   25.52   25.52   25.52   25.52   25.52   25.52   25.52   25.52
   25.52   25.52   25.52   25.52   25.52   25.52   25.52   25.52   25.52   25.52
   25.52   25.52   25.52   25.52   25.52   25.52   25.52   25.52   25.52   25.52
   25.52   25.52   25.52   25.52   25.52   25.52   25.52   25.52   25.52   25.52
   25.52   25.52   25.52   25.52   25.52   25.52   25.52   25.52   25.52   25.52
   25.52   25.52   25.52   25.52   25.52   25.52   25.52   25.52   25.52   25.52
   25.52   25.52   25.52   25.52   25.52   25.52   25.52   25.52   25.52   25.52
   25.52   25.52   25.52   25.52   25.52   25.52   25.52   25.52   25.52   25.52
   25.52   25.52   25.52   25.52   25.52   25.52   25.52   25.52   25.52   25.52
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Use DSS=False
CWMS InputPosition= 0
Use Fixed Start Time=False
Is Critical Boundary=False
Boundary Location=Churchill River ,Main            ,9566.389,        ,                ,                ,
Interval=1HOUR
Lateral Inflow Hydrograph= 744
  290.88  290.88  290.88  290.88  290.88  290.88  290.88  290.88  290.88  290.88
  290.88  290.88  290.88  290.88  290.88  290.88  290.88  290.88  290.88  290.88
  290.88  290.88  290.88  290.88  290.88  290.88  290.88  290.88  290.88  290.88
  290.88  290.88  290.88  290.88  290.88  290.88  290.88  290.88  290.88  290.88
  290.88  290.88  290.88  290.88  290.88  290.88  290.88  290.88  290.88  290.88
  290.88  290.88  290.88  290.88  290.88  290.88  290.88  290.88  290.88  290.88
  290.88  290.88  290.88  290.88  290.88  290.88  290.88  290.88  290.88  290.88
  290.88  290.88  290.88  290.88  290.88  290.88  290.88  290.88  290.88  290.88
  290.88  290.88  290.88  290.88  290.88  290.88  290.88  290.88  290.88  290.88
  290.88  290.88  290.88  290.88  290.88  290.88  290.88  290.88  290.88  290.88
  290.88  290.88  290.88  290.88  290.88  290.88  290.88  290.88  290.88  290.88
  290.88  290.88  290.88  290.88  290.88  290.88  290.88  290.88  290.88  290.88
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Use DSS=False
CWMS InputPosition= 0
Use Fixed Start Time=False
Is Critical Boundary=False
Boundary Location=Churchill River ,Main DS         ,-1972.08,        ,                ,                ,
Interval=1HOUR
Stage Hydrograph= 744
     .22     .22     .22     .22     .22     .22     .22     .22     .22     .22
     .22     .22     .22     .22     .22     .22     .22     .22     .22     .22
     .22     .22     .22     .22     .22     .22     .22     .22     .22     .22
     .22     .22     .22     .22     .22     .22     .22     .22     .22     .22
     .22     .22     .22     .22     .22     .22     .22     .22     .22     .22
     .22     .22     .22     .22     .22     .22     .22     .22     .22     .22
     .22     .22     .22     .22     .22     .22     .22     .22     .22     .22
     .22     .22     .22     .22     .22     .22     .22     .22     .22     .22
     .22     .22     .22     .22     .22     .22     .22     .22     .22     .22
     .22     .22     .22     .22     .22     .22     .22     .22     .22     .22
     .22     .22     .22     .22     .22     .22     .22     .22     .22     .22
     .22     .22     .22     .22     .22     .22     .22     .22     .22     .22
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Use DSS=False
CWMS InputPosition= 0
Use Fixed Start Time=False
Is Critical Boundary=False
