HEC-RAS study Churchill_Mapping.prj: Churchill River Flood Risk Mapping

--- Churchill_Mapping.u10 (unsteady flow) ---

Flow Title=20 Year CC
Program Version=4.10
Use Restart= 0
Initial Flow Loc=Churchill River ,Main            ,41243.44,1508
Initial Flow Loc=Churchill River ,Main DS         ,874.7763,1511.4
Initial Flow Loc=Mud Lake A      ,Main A          ,4343.607,1.7
Initial Flow Loc=Mud Lake B      ,Main            ,5538.203,1.7
Initial Flow Loc=Mud Lake C      ,Main            ,3296.746,3.4
Initial Flow Loc=Mud Lake C      ,Main            ,2548.565,3.4
Initial Flow Loc=Mud Lake In     ,In              ,100     ,3.4
Initial Storage Elev=Mud Lake        ,0.5
Boundary Location=Churchill River ,Main            ,41243.44,        ,                ,                ,
Interval=1HOUR
Flow Hydrograph= 744
    5920    5920    5920    5920    5920    5920    5920    5920    5920    5920
    5920    5920    5920    5920    5920    5920    5920    5920    5920    5920
    5920    5920    5920    5920    5920    5920    5920    5920    5920    5920
    5920    5920    5920    5920    5920    5920    5920    5920    5920    5920
    5920    5920    5920    5920    5920    5920    5920    5920    5920    5920
    5920    5920    5920    5920    5920    5920    5920    5920    5920    5920
    5920    5920    5920    5920    5920    5920    5920    5920    5920    5920
    5920    5920    5920    5920    5920    5920    5920    5920    5920    5920
    5920    5920    5920    5920    5920    5920    5920    5920    5920    5920
    5920    5920    5920    5920    5920    5920    5920    5920    5920    5920
    5920    5920    5920    5920    5920    5920    5920    5920    5920    5920
    5920    5920    5920    5920    5920    5920    5920    5920    5920    5920
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Use DSS=False
CWMS InputPosition= 0
Use Fixed Start Time=False
Is Critical Boundary=False
Boundary Location=Mud Lake In     ,In              ,100     ,        ,                ,                ,
Interval=1HOUR
Flow Hydrograph= 767
   39.69   39.69   39.69   39.69   39.69   39.69   39.69   39.69   39.69   39.69
   39.69   39.69   39.69   39.69   39.69   39.69   39.69   39.69   39.69   39.69
   39.69   39.69   39.69   39.69   39.69   39.69   39.69   39.69   39.69   39.69
   39.69   39.69   39.69   39.69   39.69   39.69   39.69   39.69   39.69   39.69
   39.69   39.69   39.69   39.69   39.69   39.69   39.69   39.69   39.69   39.69
   39.69   39.69   39.69   39.69   39.69   39.69   39.69   39.69   39.69   39.69
   39.69   39.69   39.69   39.69   39.69   39.69   39.69   39.69   39.69   39.69
   39.69   39.69   39.69   39.69   39.69   39.69   39.69   39.69   39.69   39.69
   39.69   39.69   39.69   39.69   39.69   39.69   39.69   39.69   39.69   39.69
   39.69   39.69   39.69   39.69   39.69   39.69   39.69   39.69   39.69   39.69
   39.69   39.69   39.69   39.69   39.69   39.69   39.69   39.69   39.69   39.69
   39.69   39.69   39.69   39.69   39.69   39.69   39.69   39.69   39.69   39.69
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Use DSS=False
CWMS InputPosition= 0
Use Fixed Start Time=False
Is Critical Boundary=False
Boundary Location=Churchill River ,Main            ,40242.1 ,        ,                ,                ,
Interval=1HOUR
Lateral Inflow Hydrograph= 744
   65.67   65.67   65.67   65.67   65.67   65.67   65.67   65.67   65.67   65.67
   65.67   65.67   65.67   65.67   65.67   65.67   65.67   65.67   65.67   65.67
   65.67   65.67   65.67   65.67   65.67   65.67   65.67   65.67   65.67   65.67
   65.67   65.67   65.67   65.67   65.67   65.67   65.67   65.67   65.67   65.67
   65.67   65.67   65.67   65.67   65.67   65.67   65.67   65.67   65.67   65.67
   65.67   65.67   65.67   65.67   65.67   65.67   65.67   65.67   65.67   65.67
   65.67   65.67   65.67   65.67   65.67   65.67   65.67   65.67   65.67   65.67
   65.67   65.67   65.67   65.67   65.67   65.67   65.67   65.67   65.67   65.67
   65.67   65.67   65.67   65.67   65.67   65.67   65.67   65.67   65.67   65.67
   65.67   65.67   65.67   65.67   65.67   65.67   65.67   65.67   65.67   65.67
   65.67   65.67   65.67   65.67   65.67   65.67   65.67   65.67   65.67   65.67
   65.67   65.67   65.67   65.67   65.67   65.67   65.67   65.67   65.67   65.67
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Use DSS=False
CWMS InputPosition= 0
Use Fixed Start Time=False
Is Critical Boundary=False
Boundary Location=Churchill River ,Main            ,36181.25,        ,                ,                ,
Interval=1HOUR
Lateral Inflow Hydrograph= 744
   19.32   19.32   19.32   19.32   19.32   19.32   19.32   19.32   19.32   19.32
   19.32   19.32   19.32   19.32   19.32   19.32   19.32   19.32   19.32   19.32
   19.32   19.32   19.32   19.32   19.32   19.32   19.32   19.32   19.32   19.32
   19.32   19.32   19.32   19.32   19.32   19.32   19.32   19.32   19.32   19.32
   19.32   19.32   19.32   19.32   19.32   19.32   19.32   19.32   19.32   19.32
   19.32   19.32   19.32   19.32   19.32   19.32   19.32   19.32   19.32   19.32
   19.32   19.32   19.32   19.32   19.32   19.32   19.32   19.32   19.32   19.32
   19.32   19.32   19.32   19.32   19.32   19.32   19.32   19.32   19.32   19.32
   19.32   19.32   19.32   19.32   19.32   19.32   19.32   19.32   19.32   19.32
   19.32   19.32   19.32   19.32   19.32   19.32   19.32   19.32   19.32   19.32
   19.32   19.32   19.32   19.32   19.32   19.32   19.32   19.32   19.32   19.32
   19.32   19.32   19.32   19.32   19.32   19.32   19.32   19.32   19.32   19.32
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Use DSS=False
CWMS InputPosition= 0
Use Fixed Start Time=False
Is Critical Boundary=False
Boundary Location=Churchill River ,Main            ,25199.9 ,        ,                ,                ,
Interval=1HOUR
Lateral Inflow Hydrograph= 744
   28.16   28.16   28.16   28.16   28.16   28.16   28.16   28.16   28.16   28.16
   28.16   28.16   28.16   28.16   28.16   28.16   28.16   28.16   28.16   28.16
   28.16   28.16   28.16   28.16   28.16   28.16   28.16   28.16   28.16   28.16
   28.16   28.16   28.16   28.16   28.16   28.16   28.16   28.16   28.16   28.16
   28.16   28.16   28.16   28.16   28.16   28.16   28.16   28.16   28.16   28.16
   28.16   28.16   28.16   28.16   28.16   28.16   28.16   28.16   28.16   28.16
   28.16   28.16   28.16   28.16   28.16   28.16   28.16   28.16   28.16   28.16
   28.16   28.16   28.16   28.16   28.16   28.16   28.16   28.16   28.16   28.16
   28.16   28.16   28.16   28.16   28.16   28.16   28.16   28.16   28.16   28.16
   28.16   28.16   28.16   28.16   28.16   28.16   28.16   28.16   28.16   28.16
   28.16   28.16   28.16   28.16   28.16   28.16   28.16   28.16   28.16   28.16
   28.16   28.16   28.16   28.16   28.16   28.16   28.16   28.16   28.16   28.16
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Use DSS=False
CWMS InputPosition= 0
Use Fixed Start Time=False
Is Critical Boundary=False
Boundary Location=Churchill River ,Main            ,13613.57,        ,                ,                ,
Interval=1HOUR
Lateral Inflow Hydrograph= 744
   21.59   21.59   21.59   21.59   21.59   21.59   21.59   21.59   21.59   21.59
   21.59   21.59   21.59   21.59   21.59   21.59   21.59   21.59   21.59   21.59
   21.59   21.59   21.59   21.59   21.59   21.59   21.59   21.59   21.59   21.59
   21.59   21.59   21.59   21.59   21.59   21.59   21.59   21.59   21.59   21.59
   21.59   21.59   21.59   21.59   21.59   21.59   21.59   21.59   21.59   21.59
   21.59   21.59   21.59   21.59   21.59   21.59   21.59   21.59   21.59   21.59
   21.59   21.59   21.59   21.59   21.59   21.59   21.59   21.59   21.59   21.59
   21.59   21.59   21.59   21.59   21.59   21.59   21.59   21.59   21.59   21.59
   21.59   21.59   21.59   21.59   21.59   21.59   21.59   21.59   21.59   21.59
   21.59   21.59   21.59   21.59   21.59   21.59   21.59   21.59   21.59   21.59
   21.59   21.59   21.59   21.59   21.59   21.59   21.59   21.59   21.59   21.59
   21.59   21.59   21.59   21.59   21.59   21.59   21.59   21.59   21.59   21.59
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Use DSS=False
CWMS InputPosition= 0
Use Fixed Start Time=False
Is Critical Boundary=False
Boundary Location=Churchill River ,Main            ,9566.389,        ,                ,                ,
Interval=1HOUR
Lateral Inflow Hydrograph= 744
  247.42  247.42  247.42  247.42  247.42  247.42  247.42  247.42  247.42  247.42
  247.42  247.42  247.42  247.42  247.42  247.42  247.42  247.42  247.42  247.42
  247.42  247.42  247.42  247.42  247.42  247.42  247.42  247.42  247.42  247.42
  247.42  247.42  247.42  247.42  247.42  247.42  247.42  247.42  247.42  247.42
  247.42  247.42  247.42  247.42  247.42  247.42  247.42  247.42  247.42  247.42
  247.42  247.42  247.42  247.42  247.42  247.42  247.42  247.42  247.42  247.42
  247.42  247.42  247.42  247.42  247.42  247.42  247.42  247.42  247.42  247.42
  247.42  247.42  247.42  247.42  247.42  247.42  247.42  247.42  247.42  247.42
  247.42  247.42  247.42  247.42  247.42  247.42  247.42  247.42  247.42  247.42
  247.42  247.42  247.42  247.42  247.42  247.42  247.42  247.42  247.42  247.42
  247.42  247.42  247.42  247.42  247.42  247.42  247.42  247.42  247.42  247.42
  247.42  247.42  247.42  247.42  247.42  247.42  247.42  247.42  247.42  247.42
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Use DSS=False
CWMS InputPosition= 0
Use Fixed Start Time=False
Is Critical Boundary=False
Boundary Location=Churchill River ,Main DS         ,-1972.08,        ,                ,                ,
Interval=1HOUR
Stage Hydrograph= 744
     .22     .22     .22     .22     .22     .22     .22     .22     .22     .22
     .22     .22     .22     .22     .22     .22     .22     .22     .22     .22
     .22     .22     .22     .22     .22     .22     .22     .22     .22     .22
     .22     .22     .22     .22     .22     .22     .22     .22     .22     .22
     .22     .22     .22     .22     .22     .22     .22     .22     .22     .22
     .22     .22     .22     .22     .22     .22     .22     .22     .22     .22
     .22     .22     .22     .22     .22     .22     .22     .22     .22     .22
     .22     .22     .22     .22     .22     .22     .22     .22     .22     .22
     .22     .22     .22     .22     .22     .22     .22     .22     .22     .22
     .22     .22     .22     .22     .22     .22     .22     .22     .22     .22
     .22     .22     .22     .22     .22     .22     .22     .22     .22     .22
     .22     .22     .22     .22     .22     .22     .22     .22     .22     .22
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Use DSS=False
CWMS InputPosition= 0
Use Fixed Start Time=False
Is Critical Boundary=False

--- Churchill_Mapping.u13 (unsteady flow) ---

Flow Title=2018 Jun - Aug Clipped
Program Version=4.10
Use Restart= 0
Initial Flow Loc=Churchill River ,Main            ,41243.44,3785
Initial Flow Loc=Churchill River ,Main DS         ,874.7763,3800.2
Initial Flow Loc=Mud Lake A      ,Main A          ,4343.607,7.6
Initial Flow Loc=Mud Lake B      ,Main            ,5538.203,7.6
Initial Flow Loc=Mud Lake C      ,Main            ,3296.746,7.6
Initial Flow Loc=Mud Lake C      ,Main            ,2548.565,15.2
Initial Flow Loc=Mud Lake In     ,In              ,100     ,15.2
Initial Storage Elev=Mud Lake        ,0.5
Boundary Location=Churchill River ,Main            ,41243.44,        ,                ,                ,
Interval=1HOUR
Flow Hydrograph= 1464
3785.4953784.7843786.4073788.1633788.2973789.1953790.6283793.211 3793.843796.502
4062.073 4052.46 4052.434053.3744054.375 4051.344052.2834172.9424172.6184172.556
4172.8494169.3094173.5294174.889 4320.684324.4854325.849 4328.354331.2034336.247
4518.1644522.8344527.735 4861.824834.1724834.5894837.2894844.1584840.5024843.471
4847.7894999.2415006.7425014.9725020.9335023.9935024.8135027.3055078.4635082.915
5080.8165086.5415083.138  5086.75087.0825087.4635087.5595095.0045087.2415089.754
 5091.445085.937 5087.055084.8555082.7565081.2295079.2585081.3564943.4724950.209
4948.3694951.0834953.5474949.616 4950.244952.6114949.7414950.646 4955.174944.251
4942.8174936.8614931.4064928.9434924.7064925.5164639.7574662.5664663.9634663.797
4667.349 4669.224671.1144667.3494668.675 4666.974668.8884666.3074666.4024664.981
4662.2344658.7534658.3514655.0594650.5354648.2614426.744 4440.374444.2284440.438
4446.7314444.0024445.5134441.1824443.528 4439.314441.0474439.6254302.4464312.324
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Use DSS=False
CWMS InputPosition= 0
Use Fixed Start Time=False
Is Critical Boundary=False
Boundary Location=Churchill River ,Main DS         ,32.94778,        ,                ,                ,
Interval=1HOUR
Stage Hydrograph= 1464
    .307     .36     .36    .333    .286    .245    .212.1670001    .159    .144
    .143    .194.2549999    .299    .313    .314    .302    .266    .245    .215
.2380001     .26.3149999    .377    .446.5429999    .576    .572.5470001    .524
    .472    .452    .413    .386    .371    .396    .423    .448    .488    .513
    .502    .484.4649999    .449    .443    .433    .444    .486.5419999    .601
    .622    .637     .65.5920001    .581.5669999.5519999    .507    .488      .5
    .501    .506    .553    .565    .573    .577     .56    .543.5140001.5089999
.4800001    .492    .504    .548.6019999    .602    .611    .578    .539.5000001
    .488     .45    .463    .436.4270001    .471    .469    .485     .51    .514
    .516    .489    .456    .428    .418    .394.3980001    .443    .501     .55
    .566    .534    .531    .494    .471    .439    .409    .388    .374    .361
.4029999    .412    .445    .443    .447    .446     .44    .418    .395    .385
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Use DSS=False
CWMS InputPosition= 0
Use Fixed Start Time=False
Is Critical Boundary=False
Boundary Location=Mud Lake In     ,In              ,100     ,        ,                ,                ,
Interval=1HOUR
Flow Hydrograph= 1464
    15.2    15.2    15.3    15.3    15.3    15.4    15.4    15.4    15.4    15.5
    15.5    15.5    15.6    15.6    15.6    15.6    15.7    15.7    15.7    15.8
    15.8    15.8    15.8    15.9    15.9    15.9      16      16      16    16.1
    16.1    16.1    16.1    16.2    16.2    16.2    16.3    16.3    16.3    16.4
    16.4    16.4    16.4    16.5    16.5    16.5    16.6    16.6    16.6    16.7
    16.7    16.7    16.8    16.8    16.8    16.8    16.9    16.9    16.9      17
      17      17    17.1    17.1    17.1    17.2    17.2    17.2    17.3    17.3
    17.3    17.3    17.4    17.4    17.4    17.5    17.5    17.5    17.6    17.6
    17.6    17.7    17.7    17.7    17.7    17.8    17.8    17.8    17.9    17.9
    17.9      18      18      18      18    18.1    18.1    18.1    18.2    18.2
    18.2    18.2    18.3    18.3    18.3    18.4    18.4    18.4    18.4    18.5
    18.5    18.5    18.5    18.6    18.6    18.6    18.6    18.7    18.7    18.7
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Use DSS=False
CWMS InputPosition= 0
Use Fixed Start Time=False
Is Critical Boundary=False
Boundary Location=Churchill River ,Main            ,9566.389,        ,                ,                ,
Interval=1HOUR
Lateral Inflow Hydrograph= 1464
   338.3   342.1   345.9   349.9   353.9   358.1   362.3   366.6   370.9   375.3
   379.7   384.1   388.6     393   397.4   401.8   406.1   410.3   414.4   418.4
   422.4   426.2     430   433.7   437.3   440.8   444.2   447.3   450.2   452.9
   455.3   457.5   459.4     461   462.3   463.4   464.1   464.5   464.7   464.6
   464.1   463.4   462.5   461.3   459.8     458     456   453.8   451.3   448.5
   445.5   442.3   438.9   435.2   431.4   427.4   423.3     419   414.7   410.2
   405.6   400.9   396.2   391.5   386.7   381.9     377   372.2   367.3   362.3
   357.4   352.6   347.8     343   338.5     334   329.7   325.5   321.4   317.5
   313.6   309.9   306.3   302.9   299.5   296.3   293.1   290.1   287.1   284.3
   281.6   278.9   276.2   273.7   271.1   268.6   266.1   263.7   261.3   258.8
   256.4     254   251.6   249.2   246.8   244.4   241.9   239.5     237   234.5
   231.9   229.4   226.7   224.1   221.3   218.6   215.8   212.9     210   207.1
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Use DSS=False
CWMS InputPosition= 0
Use Fixed Start Time=False
Is Critical Boundary=False
Boundary Location=Churchill River ,Main            ,40242.1 ,        ,                ,                ,
Interval=1HOUR
Lateral Inflow Hydrograph= 1464
    75.8    76.8    77.8    78.8    79.9    80.9    81.9      83      84      85
      86      87      88    88.9    89.8    90.7    91.6    92.4    93.1    93.9
    94.5    95.2    95.8    96.3    96.9    97.4    97.9    98.3    98.6    98.9
    99.1    99.3    99.4    99.4    99.3    99.2      99    98.7    98.3    97.9
    97.4    96.9    96.2    95.5    94.8    93.9    93.1    92.1    91.2    90.2
    89.2    88.1      87    85.9    84.8    83.6    82.5    81.3    80.1    78.9
    77.8    76.7    75.6    74.5    73.5    72.5    71.5    70.5    69.6    68.7
    67.9      67    66.2    65.4    64.6    63.9    63.2    62.5    61.8    61.1
    60.5    59.8    59.2    58.6    58.1    57.5      57    56.5      56    55.6
    55.1    54.7    54.3    53.9    53.5      53    52.6    52.2    51.8    51.3
    50.9    50.4    49.9    49.4    48.9    48.4    47.9    47.3    46.7    46.1
    45.5    44.9    44.2    43.6    42.9    42.2    41.5    40.8    40.1    39.4
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Use DSS=False
CWMS InputPosition= 0
Use Fixed Start Time=False
Is Critical Boundary=False
Boundary Location=Churchill River ,Main            ,36181.25,        ,                ,                ,
Interval=1HOUR
Lateral Inflow Hydrograph= 1465
    50.4    50.5    50.6    50.6    50.6    50.5    50.5    50.4    50.2    50.1
    49.9    49.8    49.6    49.4      49    48.6    48.1    47.4    46.7    45.9
    45.2    44.6    44.3    44.2    44.4    44.6    44.7    44.5    43.8    42.7
    41.1    39.3    37.4    35.6    33.9    32.4      31    29.8    28.7    27.7
    26.9    26.3    25.8    25.4      25      25      25    24.9    24.9    24.9
    24.9    24.9    24.8    24.8    24.8    24.8    24.8    24.7    24.7    24.7
    24.7    24.6    24.6    24.6    24.6    24.6    24.7    24.7    24.8    24.8
    24.9      25    25.1    25.2    25.4    25.5    25.6    25.7    25.8    25.9
      26    26.1    26.2    26.3    26.3    26.4    26.5    26.6    26.8    26.9
      27      27    26.9    26.5      26    25.4      25      25    24.9    24.9
    24.9    24.9    24.9    24.8    24.8    24.8    24.8    24.8    24.7    24.7
    24.7    24.7    24.7    24.6    24.6    24.6    24.6    24.6    24.5    24.5
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Use DSS=False
CWMS InputPosition= 0
Use Fixed Start Time=False
Is Critical Boundary=False
Boundary Location=Churchill River ,Main            ,25199.9 ,        ,                ,                ,
Interval=1HOUR
Lateral Inflow Hydrograph= 1465
    52.6    52.9    53.1    53.3    53.4    53.5    53.5    53.5    53.4    53.3
    53.2    53.1    52.9    52.7    52.3    51.9    51.3    50.5    49.7    48.7
    47.8    46.9    46.3      46      46    46.1    46.1    45.9    45.2      44
    42.3    40.3    37.9    35.4      33    30.8    28.7    26.7      25    23.4
      22    20.8    19.8      19    18.2    17.7    17.2    16.7    16.4    16.1
    15.8    15.6    15.4    15.2    15.1    14.9    14.7    14.6    14.4    14.3
    14.2    14.1      14    13.9    13.8    13.8    13.8    13.8    13.9      14
    14.1    14.2    14.3    14.5    14.6    14.8    14.9    15.1    15.2    15.4
    15.5    15.6    15.8    15.9    16.1    16.3    16.4    16.6    16.8    17.1
    17.2    17.3    17.2    16.9    16.5    15.8      15    14.1    13.2    12.3
    11.5    10.8    10.2     9.6     9.1     8.6     8.2     7.8     7.5     7.1
     6.9     6.6     6.4     6.2     6.2     6.2     6.2     6.2     6.2     6.2
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Use DSS=False
CWMS InputPosition= 0
Use Fixed Start Time=False
Is Critical Boundary=False
Boundary Location=Churchill River ,Main            ,13613.57,        ,                ,                ,
Interval=1HOUR
Lateral Inflow Hydrograph= 1465
    40.9      41    41.1    41.2    41.2    41.1      41    40.9    40.8    40.7
    40.5    40.3    40.1    39.9    39.5    39.1    38.5    37.8    36.9    36.1
    35.2    34.6    34.3    34.2    34.4    34.7    34.8    34.5    33.8    32.5
    30.7    28.7    26.5    24.5    22.6    20.9    19.3    17.9    16.6    15.6
    14.7      14    13.4    12.9    12.6    12.3    12.1      12    11.8    11.8
    11.7    11.7    11.6    11.6    11.5    11.5    11.4    11.4    11.3    11.2
    11.2    11.1    11.1    11.1    11.1    11.2    11.2    11.3    11.4    11.5
    11.6    11.7    11.8      12    12.1    12.3    12.4    12.5    12.7    12.8
    12.9      13    13.1    13.3    13.4    13.5    13.6    13.8    13.9    14.1
    14.3    14.3    14.1    13.7    13.1    12.4    11.6    10.8      10     9.4
     8.8     8.3     7.8     7.4       7     6.7     6.5     6.5     6.5     6.5
     6.5     6.5     6.5     6.5     6.5     6.4     6.4     6.4     6.4     6.4
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Use DSS=False
CWMS InputPosition= 0
Use Fixed Start Time=False
Is Critical Boundary=False

--- Churchill_Mapping.u14 (unsteady flow) ---

Flow Title=2017 Jun - Aug Clipped
Program Version=4.10
Use Restart= 0
Initial Flow Loc=Churchill River ,Main            ,41243.44,1458
Initial Flow Loc=Churchill River ,Main DS         ,874.7763,1464.2
Initial Flow Loc=Mud Lake A      ,Main A          ,4343.607,2.6
Initial Flow Loc=Mud Lake B      ,Main            ,5538.203,2.6
Initial Flow Loc=Mud Lake C      ,Main            ,3296.746,2.6
Initial Flow Loc=Mud Lake C      ,Main            ,2548.565,6.2
Initial Flow Loc=Mud Lake In     ,In              ,100     ,6.2
Initial Storage Elev=Mud Lake        ,0.5
Boundary Location=Churchill River ,Main            ,41243.44,        ,                ,                ,
Interval=1HOUR
Flow Hydrograph= 2209
1458.3451459.2141459.2141459.2141459.2141459.2141459.2141459.2141459.2141459.214
1459.2141459.2141459.2141569.3841569.3841569.3841569.3841569.3841569.3841569.384
1569.3841569.3841569.3841569.3841569.3841569.1071569.1071569.1071569.1071569.107
1569.1071569.1071569.1071569.1071569.1071569.1071569.1071588.6281588.6281588.628
1588.6281588.6281588.6281588.6281588.6281588.6281588.6281588.6281588.6281589.781
1589.7811589.7811589.7811589.7811589.7811589.7811589.7811589.7811589.7811589.781
1589.7811589.7811685.0821685.0821685.0821685.0821685.0821685.0821685.0821685.082
1685.0821685.0821685.0821682.4451682.4451682.4451682.4451682.4451682.4451682.445
1682.4451682.4451682.4451682.445 1616.28 1616.28 1616.28 1616.28 1616.28 1616.28
 1616.28 1616.28 1616.28 1616.28 1616.28 1616.28 1616.281617.9541617.9541617.954
1617.9541617.9541617.9541617.9541617.9541617.9541617.9541617.9541617.9541617.954
1617.9541617.9541617.9541617.9541617.9541617.9541617.9541617.9541617.9541617.954
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Use DSS=False
CWMS InputPosition= 0
Use Fixed Start Time=False
Is Critical Boundary=False
Boundary Location=Churchill River ,Main DS         ,32.94778,        ,                ,                ,
Interval=1HOUR
Stage Hydrograph= 2209
   -.023    .075    .152    .173     .16    .119    .056   -.015   -.082   -.147
   -.199   -.227   -.236    -.19    -.13   -.077   -.041   -.055   -.091   -.137
   -.188   -.232    -.25   -.255   -.227   -.168   -.091    -.02    .015    .008
   -.036   -.097    -.16   -.221   -.279   -.317   -.343   -.336   -.283   -.204
   -.151   -.117   -.121   -.155   -.202   -.243   -.269   -.288   -.281   -.246
   -.176   -.109   -.048   -.025   -.034    -.07   -.125   -.185    -.24   -.293
   -.337   -.349   -.337   -.288   -.214   -.145   -.107   -.102   -.142   -.187
   -.222   -.253    -.26   -.265    -.24    -.19   -.107   -.058   -.036   -.048
   -.082   -.124   -.181   -.229   -.267   -.304   -.306   -.281   -.205   -.128
   -.061   -.019   -.012   -.029   -.071   -.111   -.143   -.169   -.175   -.159
   -.109   -.028    .041    .084    .089    .055   -.001   -.048   -.093   -.134
   -.162   -.147   -.105   -.038    .065    .138    .186    .201     .18    .124
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Use DSS=False
CWMS InputPosition= 0
Use Fixed Start Time=False
Is Critical Boundary=False
Boundary Location=Mud Lake In     ,In              ,100     ,        ,                ,                ,
Interval=1HOUR
Flow Hydrograph= 2209
     6.2     6.2     6.2     6.2     6.2     6.2     6.2     6.2     6.2     6.2
     6.2     6.2     6.2     6.2     6.2     6.2     6.2     6.2     6.2     6.2
     6.1     6.1     6.1     6.1     6.1     6.1     6.1     6.1     6.1     6.1
     6.1     6.1     6.1     6.1     6.1     6.1     6.1     6.1     6.1       6
       6       6       6       6       6       6       6       6       6       6
       6       6       6       6       6       6       6       6       6     5.9
     5.9     5.9     5.9     5.9     5.9     5.9     5.9     5.9     5.9     5.9
     5.9     5.9     5.9     5.9     5.9     5.9     5.9     5.9     5.9     5.8
     5.8     5.8     5.8     5.8     5.8     5.8     5.8     5.8     5.8     5.8
     5.8     5.8     5.8     5.8     5.8     5.8     5.8     5.8     5.8     5.8
     5.7     5.7     5.7     5.7     5.7     5.7     5.7     5.7     5.7     5.7
     5.7     5.7     5.7     5.7     5.7     5.7     5.7     5.7     5.7     5.7
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Use DSS=False
CWMS InputPosition= 0
Use Fixed Start Time=False
Is Critical Boundary=False
Boundary Location=Churchill River ,Main            ,40242.1 ,        ,                ,                ,
Interval=1HOUR
Lateral Inflow Hydrograph= 2209
    17.4    17.5    17.6    17.6    17.6    17.6    17.6    17.5    17.4    17.3
    17.1      17    16.8    16.6    16.5    16.3    16.1    15.9    15.7    15.5
    15.4    15.2      15    14.9    14.7    14.6    14.4    14.3    14.2      14
    13.9    13.8    13.7    13.6    13.5    13.4    13.3    13.2    13.1      13
    12.9    12.8    12.7    12.6    12.5    12.4    12.3    12.2    12.1    11.9
    11.8    11.7    11.6    11.5    11.4    11.3    11.2    11.1    10.9    10.8
    10.7    10.6    10.5    10.4    10.3    10.2    10.1      10     9.9     9.8
     9.7     9.6     9.5     9.5     9.4     9.3     9.2     9.1       9       9
     8.9     8.8     8.7     8.7     8.6     8.5     8.5     8.4     8.3     8.3
     8.2     8.2     8.1       8       8     7.9     7.9     7.8     7.8     7.8
     7.8     7.7     7.7     7.7     7.7     7.7     7.7     7.7     7.7     7.7
     7.7     7.7     7.8     7.9       8     8.2     8.4     8.6     8.9     9.2
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Use DSS=False
CWMS InputPosition= 0
Use Fixed Start Time=False
Is Critical Boundary=False
Boundary Location=Churchill River ,Main            ,36181.25,        ,                ,                ,
Interval=1HOUR
Lateral Inflow Hydrograph= 2209
    25.2      25      25      25    24.9    24.9    24.9    24.9    24.9    24.8
    24.8    24.8    24.8    24.7    24.7    24.7    24.7    24.7    24.8    24.8
    24.9      25      25      25    25.1    25.1    25.1    25.1    25.1      25
      25      25    24.9    24.9    24.9    24.9    24.9    24.8    24.8    24.8
    24.8    24.7    24.7    24.7    24.7    24.7    24.6    24.6    24.6    24.6
    24.6    24.5    24.5    24.5    24.5    24.5    24.4    24.4    24.4    24.4
    24.4    24.3    24.3    24.3    24.3    24.3    24.2    24.2    24.2    24.2
    24.2    24.1    24.1    24.1    24.1    24.1      24      24      24      24
    23.9    23.9    23.9    23.9    23.9    23.8    23.8    23.8    23.8    23.8
    23.7    23.7    23.7    23.7    23.7    23.7    23.8    23.9    24.1    24.2
    24.4    24.4    24.5    24.5    24.4    24.4    24.4    24.4    24.4    24.3
    24.5    24.9    25.7    26.7      28    29.4    30.8    31.9    32.8    33.4
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Use DSS=False
CWMS InputPosition= 0
Use Fixed Start Time=False
Is Critical Boundary=False
Boundary Location=Churchill River ,Main            ,25199.9 ,        ,                ,                ,
Interval=1HOUR
Lateral Inflow Hydrograph= 2209
     8.7     8.4     8.1     7.9     7.7     7.5     7.3     7.1       7     6.9
     6.7     6.6     6.5     6.5     6.4     6.4     6.3     6.4     6.4     6.5
     6.6     6.6     6.7     6.8     6.9     6.9     6.9     6.9     6.9     6.9
     6.8     6.7     6.6     6.5     6.4     6.3     6.2     6.2     6.2     6.2
     6.2     6.2     6.2     6.2     6.2     6.2     6.2     6.2     6.2     6.2
     6.2     6.2     6.2     6.2     6.2     6.1     6.1     6.1     6.1     6.1
     6.1     6.1     6.1     6.1     6.1     6.1     6.1     6.1     6.1     6.1
     6.1     6.1     6.1     6.1     6.1       6       6       6       6       6
       6       6       6       6       6       6       6       6       6       6
       6       6       6       6       6       6     6.1     6.3     6.5     6.7
     6.9       7     7.1     7.2     7.2     7.1       7     6.9     6.8     6.8
     6.9     7.4     8.2     9.3    10.8    12.5    14.3      16    17.5    18.6
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Use DSS=False
CWMS InputPosition= 0
Use Fixed Start Time=False
Is Critical Boundary=False
Boundary Location=Churchill River ,Main            ,13613.57,        ,                ,                ,
Interval=1HOUR
Lateral Inflow Hydrograph= 2209
     7.7     7.5     7.3     7.2     7.1     6.9     6.8     6.7     6.7     6.6
     6.5     6.5     6.5     6.5     6.5     6.5     6.5     6.5     6.6     6.7
     6.8     6.9     6.9       7     7.1     7.1     7.1     7.2     7.1     7.1
       7     6.9     6.8     6.7     6.6     6.6     6.5     6.5     6.5     6.5
     6.5     6.5     6.5     6.5     6.5     6.4     6.4     6.4     6.4     6.4
     6.4     6.4     6.4     6.4     6.4     6.4     6.4     6.4     6.4     6.4
     6.4     6.4     6.4     6.4     6.3     6.3     6.3     6.3     6.3     6.3
     6.3     6.3     6.3     6.3     6.3     6.3     6.3     6.3     6.3     6.3
     6.3     6.3     6.3     6.2     6.2     6.2     6.2     6.2     6.2     6.2
     6.2     6.2     6.2     6.2     6.3     6.3     6.4     6.5     6.7     6.9
     7.1     7.2     7.3     7.2     7.2       7     6.9     6.8     6.7     6.7
     6.9     7.5     8.3     9.5      11    12.6    14.2    15.5    16.5    17.2
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Use DSS=False
CWMS InputPosition= 0
Use Fixed Start Time=False
Is Critical Boundary=False
Boundary Location=Churchill River ,Main            ,9566.389,        ,                ,                ,
Interval=1HOUR
Lateral Inflow Hydrograph= 2209
    58.2      59    59.9    60.7    61.4    62.1    62.7    63.2    63.7    64.1
    64.4    64.7    64.9      65    64.9    64.8    64.6    64.3    63.9    63.5
      63    62.5    61.9    61.3    60.6    59.9    59.2    58.5    57.8    57.1
    56.4    55.6    54.9    54.3    53.6    52.9    52.3    51.7    51.1    50.5
    49.9    49.4    48.8    48.3    47.7    47.2    46.7    46.2    45.7    45.2
    44.7    44.2    43.7    43.2    42.7    42.3    41.8    41.3    40.8    40.4
    39.9    39.4      39    38.5      38    37.5      37    36.6    36.1    35.6
    35.2    34.7    34.2    33.8    33.3    32.9    32.5      32    31.6    31.2
    30.8    30.4    30.1    29.7    29.3      29    28.6    28.3    27.9    27.6
    27.3      27    26.6    26.3    26.1    25.8    25.5    25.3      25    24.8
    24.6    24.4    24.2    24.1    23.9    23.8    23.6    23.5    23.4    23.3
    23.2    23.2    23.3    23.5    23.8    24.3    24.8    25.4    26.1      27
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Use DSS=False
CWMS InputPosition= 0
Use Fixed Start Time=False
Is Critical Boundary=False

--- Churchill_Mapping.u15 (unsteady flow) ---

Flow Title=2017 Oct - Nov Clipped
Program Version=4.10
Use Restart= 0
Initial Flow Loc=Churchill River ,Main            ,41243.44,1508
Initial Flow Loc=Churchill River ,Main DS         ,874.7763,1511.4
Initial Flow Loc=Mud Lake A      ,Main A          ,4343.607,1.7
Initial Flow Loc=Mud Lake B      ,Main            ,5538.203,1.7
Initial Flow Loc=Mud Lake C      ,Main            ,3296.746,1.7
Initial Flow Loc=Mud Lake C      ,Main            ,2548.565,3.4
Initial Flow Loc=Mud Lake In     ,In              ,100     ,3.4
Initial Storage Elev=Mud Lake        ,0.5
Boundary Location=Churchill River ,Main            ,41243.44,        ,                ,                ,
Interval=1HOUR
Flow Hydrograph= 744
    1508    1507    1507    1507    1507    1508    1507    1507    1507    1507
    1508    1508    1429    1429    1429    1429    1429    1429    1429    1429
    1429    1429    1430    1430    1430    1430    1430    1430    1430    1430
    1430    1431    1431    1431    1431    1431    1432    1432    1432    1432
    1432    1432    1403    1402    1403    1403    1402    1403    1403    1402
    1402    1402    1402    1402    1402    1402    1402    1402    1402    1341
    1341    1341    1342    1342    1342    1341    1342    1342    1341    1341
    1341    1341    1341    1341    1341    1341    1341    1341    1341    1340
    1340    1340    1340    1340    1309    1310    1310    1310    1310    1310
    1310    1311    1311    1311    1311    1311    1311    1311    1311    1312
    1312    1312    1312    1312    1312    1312    1312    1313    1403    1403
    1403    1403    1403    1403    1403    1403    1403    1402    1402    1402
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Use DSS=False
CWMS InputPosition= 0
Use Fixed Start Time=False
Is Critical Boundary=False
Boundary Location=Churchill River ,Main DS         ,32.94778,        ,                ,                ,
Interval=1HOUR
Stage Hydrograph= 744
   -.122    -.19   -.241   -.269   -.283   -.265   -.221   -.139   -.059    -.03
   -.048   -.096    -.16   -.203   -.234    -.26   -.252   -.227    -.15   -.039
    .061    .119    .121    .075   -.004    -.08   -.148   -.191   -.207   -.174
    -.09    .021    .135    .209     .24    .223    .154    .074    .005   -.059
   -.105   -.118   -.078    .013    .113    .199    .222    .199    .138    .056
   -.034   -.106   -.175   -.214   -.209   -.135   -.017    .087    .157    .153
    .111    .034   -.048   -.126   -.192   -.239   -.241   -.175   -.064    .051
    .121    .133    .088    .011    -.08   -.165   -.238   -.294   -.306   -.256
    -.15   -.019    .087    .131    .112    .048   -.036   -.122   -.188   -.238
   -.263   -.226   -.125    .002    .125    .189    .173    .098   -.003   -.099
    -.19   -.262    -.31   -.303    -.23   -.107    .018     .09    .112    .072
   -.003   -.092   -.186   -.256    -.31   -.323   -.273    -.18   -.069    .036
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Use DSS=False
CWMS InputPosition= 0
Use Fixed Start Time=False
Is Critical Boundary=False
Boundary Location=Mud Lake In     ,In              ,100     ,        ,                ,                ,
Interval=1HOUR
Flow Hydrograph= 767
     3.4     3.4     3.4     3.4     3.4     3.4     3.4     3.4     3.4     3.4
     3.4     3.4     3.4     3.4     3.4     3.4     3.4     3.4     3.4     3.4
     3.4     3.4     3.3     3.3     3.3     3.3     3.3     3.3     3.3     3.3
     3.3     3.3     3.3     3.3     3.3     3.3     3.3     3.3     3.3     3.3
     3.3     3.3     3.3     3.3     3.3     3.3     3.3     3.3     3.3     3.3
     3.3     3.3     3.3     3.3     3.3     3.3     3.3     3.3     3.2     3.2
     3.2     3.2     3.2     3.2     3.2     3.2     3.2     3.2     3.2     3.2
     3.2     3.2     3.2     3.2     3.2     3.2     3.2     3.2     3.2     3.2
     3.2     3.2     3.2     3.2     3.2     3.2     3.2     3.2     3.2     3.2
     3.2     3.2     3.2     3.2     3.2     3.1     3.1     3.1     3.1     3.1
     3.1     3.1     3.1     3.1     3.1     3.1     3.1     3.1     3.1     3.1
     3.1     3.1     3.1     3.1     3.1     3.1     3.1     3.1     3.1     3.1
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Use DSS=False
CWMS InputPosition= 0
Use Fixed Start Time=False
Is Critical Boundary=False
Boundary Location=Churchill River ,Main            ,40242.1 ,        ,                ,                ,
Interval=1HOUR
Lateral Inflow Hydrograph= 744
     7.2     7.2     7.3     7.3     7.4     7.4     7.5     7.5     7.6     7.6
     7.7     7.7     7.8     7.8     7.8     7.9     7.9     7.9     7.9       8
       8       8       8       8       8     7.9     7.9     7.9     7.9     7.9
     7.8     7.8     7.8     7.8     7.7     7.7     7.7     7.7     7.6     7.6
     7.6     7.6     7.6     7.6     7.6     7.6     7.6     7.6     7.6     7.6
     7.6     7.6     7.6     7.7     7.7     7.7     7.7     7.7     7.7     7.7
     7.7     7.7     7.7     7.7     7.7     7.7     7.7     7.7     7.7     7.7
     7.7     7.6     7.6     7.6     7.5     7.5     7.5     7.5     7.5     7.5
     7.5     7.5     7.5     7.5     7.4     7.4     7.4     7.4     7.4     7.4
     7.4     7.4     7.4     7.4     7.4     7.4     7.4     7.4     7.4     7.4
     7.3     7.3     7.3     7.3     7.3     7.3     7.3     7.3     7.3     7.3
     7.3     7.3     7.3     7.3     7.3     7.3     7.2     7.2     7.2     7.2
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Use DSS=False
CWMS InputPosition= 0
Use Fixed Start Time=False
Is Critical Boundary=False
Boundary Location=Churchill River ,Main            ,36181.25,        ,                ,                ,
Interval=1HOUR
Lateral Inflow Hydrograph= 744
    23.6    23.6    23.7    23.7    23.7    23.6    23.6    23.5    23.5    23.5
    23.5    23.5    23.4    23.4    23.4    23.4    23.4    23.3    23.3    23.3
    23.3    23.3    23.2    23.2    23.2    23.2    23.2    23.1    23.1    23.1
    23.1    23.1    23.1      23      23      23      23    23.1    23.1    23.2
    23.3    23.4    23.5    23.6    23.6    23.6    23.6    23.6    23.6    23.6
    23.5    23.5    23.5    23.5    23.5    23.4    23.4    23.4    23.4    23.4
    23.3    23.3    23.3    23.3    23.3    23.2    23.2    23.2    23.2    23.2
    23.1    23.1    23.1    23.1    23.1      23      23      23      23      23
    22.9    22.9    22.9    22.9    22.9    22.9    22.8    22.8    22.8    22.8
    22.8    22.8    22.7    22.7    22.7    22.7    22.7    22.7    22.7    22.6
    22.6    22.6    22.6    22.6    22.5    22.5    22.5    22.5    22.5    22.5
    22.4    22.4    22.4    22.4    22.4    22.4    22.3    22.3    22.3    22.3
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Use DSS=False
CWMS InputPosition= 0
Use Fixed Start Time=False
Is Critical Boundary=False
Boundary Location=Churchill River ,Main            ,25199.9 ,        ,                ,                ,
Interval=1HOUR
Lateral Inflow Hydrograph= 744
       7     7.1     7.2     7.2     7.3     7.3     7.2     7.1       7     6.9
     6.8     6.7     6.6     6.5     6.4     6.4     6.3     6.2     6.2     6.2
     6.2     6.2     6.2     6.2     6.2     6.2     6.2     6.2     6.2     6.2
     6.2     6.2     6.2     6.2     6.2     6.2     6.2     6.3     6.3     6.5
     6.6     6.8     6.9       7     7.1     7.2     7.2     7.2     7.1       7
     6.9     6.8     6.7     6.6     6.6     6.5     6.4     6.4     6.3     6.3
     6.2     6.2     6.2     6.2     6.2     6.2     6.2     6.2     6.2     6.2
     6.2     6.2     6.2     6.2     6.2     6.2     6.2     6.2     6.2     6.1
     6.1     6.1     6.1     6.1     6.1     6.1     6.1     6.1     6.1     6.1
     6.1     6.1     6.1     6.1     6.1     6.1     6.1     6.1     6.1     6.1
     6.1     6.1     6.1     6.1     6.1     6.1     6.1     6.1     6.1     6.1
       6       6       6       6       6       6       6       6       6       6
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Use DSS=False
CWMS InputPosition= 0
Use Fixed Start Time=False
Is Critical Boundary=False
Boundary Location=Churchill River ,Main            ,13613.57,        ,                ,                ,
Interval=1HOUR
Lateral Inflow Hydrograph= 744
       5       5     5.1     5.2     5.4     5.6     5.9     6.1     6.4     6.7
       7     7.3     7.6     7.9     8.1     8.3     8.5     8.6     8.6     8.5
     8.3     8.1     7.8     7.5     7.2     6.9     6.6     6.5     6.5     6.5
     6.5     6.5     6.5     6.5     6.5     6.5     6.4     6.4     6.4     6.4
     6.4     6.4     6.4     6.4     6.4     6.4     6.4     6.4     6.4     6.4
     6.4     6.4     6.5     6.5     6.7     6.8     6.9     7.1     7.2     7.3
     7.4     7.5     7.6     7.6     7.7     7.8     7.8     7.8     7.9     7.9
     7.9     7.9     7.9     7.9     7.9     7.9     7.9     7.9     7.9     7.9
     7.9     7.9     7.8     7.7     7.6     7.5     7.4     7.3     7.2       7
     6.9     6.8     6.7     6.6     6.5     6.5     6.5     6.5     6.5     6.5
     6.5     6.5     6.5     6.5     6.4     6.4     6.4     6.4     6.4     6.4
     6.4     6.4     6.4     6.4     6.4     6.4     6.4     6.4     6.4     6.4
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Use DSS=False
CWMS InputPosition= 0
Use Fixed Start Time=False
Is Critical Boundary=False
Boundary Location=Churchill River ,Main            ,9566.389,        ,                ,                ,
Interval=1HOUR
Lateral Inflow Hydrograph= 744
    15.6    15.7    15.8      16    16.1    16.2    16.4    16.5    16.7    16.8
      17    17.2    17.3    17.5    17.6    17.8    17.9    18.1    18.2    18.4
    18.5    18.6    18.7    18.8    18.9      19    19.1    19.2    19.2    19.3
    19.3    19.3    19.4    19.4    19.3    19.3    19.3    19.2    19.2    19.1
    19.1    19.1      19      19      19      19      19    18.9    18.9    18.9
    18.9    18.9    18.8    18.8    18.8    18.8    18.8    18.8    18.8    18.9
    18.9    18.9    18.9    18.9      19      19      19      19      19      19
      19      19    18.9    18.9    18.9    18.8    18.8    18.7    18.7    18.6
    18.6    18.5    18.4    18.3    18.2    18.1      18    17.8    17.7    17.6
    17.5    17.3    17.2    17.1      17    16.9    16.8    16.7    16.6    16.5
    16.4    16.3    16.2    16.1      16      16      16      16    15.9    15.9
    15.9    15.9    15.9    15.9    15.9    15.9    15.8    15.8    15.8    15.8
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Use DSS=False
CWMS InputPosition= 0
Use Fixed Start Time=False
Is Critical Boundary=False
