--- Churchill_Forecasting.prj (project) ---

Proj Title=ChurchillRiver_Forecasting
Current Plan=p09
Default Exp/Contr=0.3,0.1
SI Units
Geom File=g11
Geom File=g14
Flow File=f02
Unsteady File=u05
Unsteady File=u06
Unsteady File=u07
Unsteady File=u08
Unsteady File=u09
Unsteady File=u04
Plan File=p04
Plan File=p06
Plan File=p07
Plan File=p09
Plan File=p12
Plan File=p13
Plan File=p14
Y Axis Title=Elevation
X Axis Title(PF)=Main Channel Distance
X Axis Title(XS)=Station
BEGIN DESCRIPTION:
END DESCRIPTION:
DSS Start Date=01JUN2018
DSS Start Time=00:00
DSS End Date=31JUL2018
DSS End Time=23:00
DSS Export Rating Curves= 0
DSS Export Rating Curve Sorted= 0
DSS Export Volume Flow Curves= 0
DXF Filename=P:\Projects\2018\18-3217-001\Design\Hydr\Hydraulic Modelling\Open Water\HEC-RAS Model\Rev 1 Model - Nalcor LiDAR\ChurchillRiver.
DXF OffsetX= 0
DXF OffsetY= 0
DXF ScaleX= 1
DXF ScaleY= 10

--- Churchill_Forecasting.p09 (plan) ---

Plan Title=Rating Curves
Program Version=4.10
Short Identifier=Rating Curves
Simulation Date=15Oct2017,00:00,14Nov2017,00:00
Geom File=g11
Flow File=f02
Subcritical Flow
K Sum by GR= 0
Std Step Tol= 0.003
Critical Tol= 0.003
Num of Std Step Trials= 20
Max Error Tol= 0.1
Flow Tol Ratio= 0.001
Split Flow NTrial= 30
Split Flow Tol= 0.006
Split Flow Ratio= 0.02
Log Output Level= 0
Friction Slope Method= 1
Unsteady Friction Slope Method= 2
Unsteady Bridges Friction Slope Method= 1
Parabolic Critical Depth
Global Vel Dist= 0 , 0 , 0
Global Log Level= 0
CheckData=True
Encroach Param=-1 ,0,0, 0
Computation Interval=1HOUR
Output Interval=1HOUR
Run HTab= 1
Run UNet= 1
Run PostProcess= 1
Run WQNet= 0
UNET Theta= 1
UNET Theta Warmup= 1
UNET ZTol= 0.006
UNET ZSATol= 0.015
UNET MxIter= 20
UNET MaxInSteps= 0
UNET DtIC= 0
UNET DtMin= 0
UNET MaxCRTS= 20
UNET WFStab= 2
UNET SFStab= 1
UNET WFX= 1
UNET SFX= 1
UNET DSS MLevel= 4
UNET DZMax Abort= 30
UNET Convert EG Bridges= 0
UNET Use Existing IB Tables=-1
UNET Froude Reduction=False
UNET Froude Limit= 1
UNET Froude Power= 10
UNET Time Slicing=0,0, 5
UNET Junction Losses=0
Instantaneous Interval=1HOUR
DSS File=dss
Write IC File= 0
Write IC File at Sim End=0
Echo Input=False
Echo Parameters=False
Echo Output=False
Write Detailed= 0
WQ AD Non Conservative
WQ ULTIMATE=-1
WQ Max Comp Step=1HOUR
WQ Output Interval=15MIN
WQ Output Selected Increments= 0
WQ Output face flow=0
WQ Output face velocity=0
WQ Output face area=0
WQ Output face dispersion=0
WQ Output cell volume=0
WQ Output cell surface area=0
WQ Output cell continuity=0
WQ Output cumulative cell continuity=0
WQ Output face conc=0
WQ Output face dconc_dx=0
WQ Output face courant=0
WQ Output face peclet=0
WQ Output face adv mass=0
WQ Output face disp mass=0
WQ Output cell mass=0
WQ Output cell source sink temp=0
WQ Output cell source sink nsm=0
WQ Output MaxMinRange=-1
WQ Daily Max Min Mean=-1
WQ Daily Range=0
WQ Daily Time=0
WQ Create Restart=0
WQ Fixed Restart=0
WQ System Summary=0
WQ Use Fixed Temperature=0
Sorting and Armoring Iterations= 10
XS Update Threshold= 0.02
Hydraulics Update Threshold= 0.02
Energy Slope Method= 1
Volume Change Method= 0
XS Weighting Method= 0
Number of US Weighted Cross Sections= 1
Number of DS Weighted Cross Sections= 1
Upstream XS Weight=0.25
Main XS Weight=0.5
Downstream XS Weight=0.25
Number of DS XS's Weighted with US Boundary= 1
Upstream Boundary Weight= 1
Weight of XSs Associated with US Boundary= 0
Number of US XS's Weighted with DS Boundary= 1
Downstream Boundary Weight= 0.5
Weight of XSs Associated with DS Boundary= 0.5
Sediment Output Level= 4
Mass or Volume Output= 0
Output Increment Type= 1
Profile and TS Output Increment= 10
XS Output Flag= 0
XS Output Increment= 10
Disregard all LS=0
Disregard all Conn=0
Disregard all Breaches=0
Disregard all Pumps=0

--- Churchill_Forecasting.p04 (plan) ---

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Plan Title=Jun - Aug 2018
Short Identifier=Jun Aug 2018
Simulation Date=01JUN2018,00:00,31JUL2018,23:00
Geom File=g11
Flow File=u04

--- Churchill_Forecasting.p06 (plan) ---

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Plan Title=Jun - Aug 2017
Short Identifier=Jun Aug 2017
Simulation Date=15JUN2017,00:00,14Sep2017,00:00
Geom File=g11
Flow File=u05

--- Churchill_Forecasting.p07 (plan) ---

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Plan Title=Oct - Nov 2017
Short Identifier=Oct Nov 2017
Geom File=g11
Flow File=u06

--- Churchill_Forecasting.p12 (plan) ---

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Plan Title=Jun - Aug 2018 Clipped
Short Identifier=Jun Aug 2018 CL
Simulation Date=01JUN2018,00:00,31JUL2018,23:00
Geom File=g14
Flow File=u07

--- Churchill_Forecasting.p13 (plan) ---

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Plan Title=Jun - Aug 2017 Clipped
Short Identifier=Jun Aug 2017 CL
Simulation Date=15JUN2017,00:00,14Sep2017,00:00
Geom File=g14
Flow File=u08

--- Churchill_Forecasting.p14 (plan) ---

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Plan Title=Oct - Nov 2017 Clipped
Short Identifier=Oct Nov 2017 CL
Geom File=g14
Flow File=u09
