HEC-RAS study Churchill_Forecasting.prj: ChurchillRiver_Forecasting

--- Churchill_Forecasting.f02 (steady flow) ---

Flow Title=Rating Curves
Program Version=4.10
Number of Profiles= 735
Profile Names=PF 1,PF 2,PF 3,PF 4,PF 5,PF 6,PF 7,PF 8,PF 9,PF 10,PF 11,PF 12,PF 13,PF 14,PF 15,PF 16,PF 17,PF 18,PF 19,PF 20,PF 21,PF 22,PF 23,PF 24,PF 25,PF 26,PF 27,PF 28,PF 29,PF 30,PF 31,PF 32,PF 33,PF 34,PF 35,PF 36,PF 37,PF 38,PF 39,PF 40,PF 41,PF 42,PF 43,PF 44,PF 45,PF 46,PF 47,PF 48,PF 49,PF 50,PF 51,PF 52,PF 53,PF 54,PF 55,PF 56,PF 57,PF 58,PF 59,PF 60,PF 61,PF 62,PF 63,PF 64,PF 65,PF 66,PF 67,PF 68,PF 69,PF 70,PF 71,PF 72,PF 73,PF 74,PF 75,PF 76,PF 77,PF 78,PF 79,PF 80,PF 81,PF 82,PF 83,PF 84,PF 85,PF 86,PF 87,PF 88,PF 89,PF 90,PF 91,PF 92,PF 93,PF 94,PF 95,PF 96,PF 97,PF 98,PF 99,PF 100,PF 101,PF 102,PF 103,PF 104,PF 105,PF 106,PF 107,PF 108,PF 109,PF 110,PF 111,PF 112,PF 113,PF 114,PF 115,PF 116,PF 117,PF 118,PF 119,PF 120,PF 121,PF 122,PF 123,PF 124,PF 125,PF 126,PF 127,PF 128,PF 129,PF 130,PF 131,PF 132,PF 133,PF 134,PF 135,PF 136,PF 137,PF 138,PF 139,PF 140,PF 141,PF 142,PF 143,PF 144,PF 145,PF 146,PF 147,PF 148,PF 149,PF 150,PF 151,PF 152,PF 153,PF 154,PF 155,PF 156,PF 157,PF 158,PF 159,PF 160,PF 161,PF 162,PF 163,PF 164,PF 165,PF 166,PF 167,PF 168,PF 169,PF 170,PF 171,PF 172,PF 173,PF 174,PF 175,PF 176,PF 177,PF 178,PF 179,PF 180,PF 181,PF 182,PF 183,PF 184,PF 185,PF 186,PF 187,PF 188,PF 189,PF 190,PF 191,PF 192,PF 193,PF 194,PF 195,PF 196,PF 197,PF 198,PF 199,PF 200,PF 201,PF 202,PF 203,PF 204,PF 205,PF 206,PF 207,PF 208,PF 209,PF 210,PF 211,PF 212,PF 213,PF 214,PF 215,PF 216,PF 217,PF 218,PF 219,PF 220,PF 221,PF 222,PF 223,PF 224,PF 225,PF 226,PF 227,PF 228,PF 229,PF 230,PF 231,PF 232,PF 233,PF 234,PF 235,PF 236,PF 237,PF 238,PF 239,PF 240,PF 241,PF 242,PF 243,PF 244,PF 245,PF 246,PF 247,PF 248,PF 249,PF 250,PF 251,PF 252,PF 253,PF 254,PF 255,PF 256,PF 257,PF 258,PF 259,PF 260,PF 261,PF 262,PF 263,PF 264,PF 265,PF 266,PF 267,PF 268,PF 269,PF 270,PF 271,PF 272,PF 273,PF 274,PF 275,PF 276,PF 277,PF 278,PF 279,PF 280,PF 281,PF 282,PF 283,PF 284,PF 285,PF 286,PF 287,PF 288,PF 289,PF 290,PF 291,PF 292,PF 293,PF 294,PF 295,PF 296,PF 297,PF 298,PF 299,PF 300,PF 301,PF 302,PF 303,PF 304,PF 305,PF 306,PF 307,PF 308,PF 309,PF 310,PF 311,PF 312,PF 313,PF 314,PF 315,PF 316,PF 317,PF 318,PF 319,PF 320,PF 321,PF 322,PF 323,PF 324,PF 325,PF 326,PF 327,PF 328,PF 329,PF 330,PF 331,PF 332,PF 333,PF 334,PF 335,PF 336,PF 337,PF 338,PF 339,PF 340,PF 341,PF 342,PF 343,PF 344,PF 345,PF 346,PF 347,PF 348,PF 349,PF 350,PF 351,PF 352,PF 353,PF 354,PF 355,PF 356,PF 357,PF 358,PF 359,PF 360,PF 361,PF 362,PF 363,PF 364,PF 365,PF 366,PF 367,PF 368,PF 369,PF 370,PF 371,PF 372,PF 373,PF 374,PF 375,PF 376,PF 377,PF 378,PF 379,PF 380,PF 381,PF 382,PF 383,PF 384,PF 385,PF 386,PF 387,PF 388,PF 389,PF 390,PF 391,PF 392,PF 393,PF 394,PF 395,PF 396,PF 397,PF 398,PF 399,PF 400,PF 401,PF 402,PF 403,PF 404,PF 405,PF 406,PF 407,PF 408,PF 409,PF 410,PF 411,PF 412,PF 413,PF 414,PF 415,PF 416,PF 417,PF 418,PF 419,PF 420,PF 421,PF 422,PF 423,PF 424,PF 425,PF 426,PF 427,PF 428,PF 429,PF 430,PF 431,PF 432,PF 433,PF 434,PF 435,PF 436,PF 437,PF 438,PF 439,PF 440,PF 441,PF 442,PF 443,PF 444,PF 445,PF 446,PF 447,PF 448,PF 449,PF 450,PF 451,PF 452,PF 453,PF 454,PF 455,PF 456,PF 457,PF 458,PF 459,PF 460,PF 461,PF 462,PF 463,PF 464,PF 465,PF 466,PF 467,PF 468,PF 469,PF 470,PF 471,PF 472,PF 473,PF 474,PF 475,PF 476,PF 477,PF 478,PF 479,PF 480,PF 481,PF 482,PF 483,PF 484,PF 485,PF 486,PF 487,PF 488,PF 489,PF 490,PF 491,PF 492,PF 493,PF 494,PF 495,PF 496,PF 497,PF 498,PF 499,PF 500,PF 501,PF 502,PF 503,PF 504,PF 505,PF 506,PF 507,PF 508,PF 509,PF 510,PF 511,PF 512,PF 513,PF 514,PF 515,PF 516,PF 517,PF 518,PF 519,PF 520,PF 521,PF 522,PF 523,PF 524,PF 525,PF 526,PF 527,PF 528,PF 529,PF 530,PF 531,PF 532,PF 533,PF 534,PF 535,PF 536,PF 537,PF 538,PF 539,PF 540,PF 541,PF 542,PF 543,PF 544,PF 545,PF 546,PF 547,PF 548,PF 549,PF 550,PF 551,PF 552,PF 553,PF 554,PF 555,PF 556,PF 557,PF 558,PF 559,PF 560,PF 561,PF 562,PF 563,PF 564,PF 565,PF 566,PF 567,PF 568,PF 569,PF 570,PF 571,PF 572,PF 573,PF 574,PF 575,PF 576,PF 577,PF 578,PF 579,PF 580,PF 581,PF 582,PF 583,PF 584,PF 585,PF 586,PF 587,PF 588,PF 589,PF 590,PF 591,PF 592,PF 593,PF 594,PF 595,PF 596,PF 597,PF 598,PF 599,PF 600,PF 601,PF 602,PF 603,PF 604,PF 605,PF 606,PF 607,PF 608,PF 609,PF 610,PF 611,PF 612,PF 613,PF 614,PF 615,PF 616,PF 617,PF 618,PF 619,PF 620,PF 621,PF 622,PF 623,PF 624,PF 625,PF 626,PF 627,PF 628,PF 629,PF 630,PF 631,PF 632,PF 633,PF 634,PF 635,PF 636,PF 637,PF 638,PF 639,PF 640,PF 641,PF 642,PF 643,PF 644,PF 645,PF 646,PF 647,PF 648,PF 649,PF 650,PF 651,PF 652,PF 653,PF 654,PF 655,PF 656,PF 657,PF 658,PF 659,PF 660,PF 661,PF 662,PF 663,PF 664,PF 665,PF 666,PF 667,PF 668,PF 669,PF 670,PF 671,PF 672,PF 673,PF 674,PF 675,PF 676,PF 677,PF 678,PF 679,PF 680,PF 681,PF 682,PF 683,PF 684,PF 685,PF 686,PF 687,PF 688,PF 689,PF 690,PF 691,PF 692,PF 693,PF 694,PF 695,PF 696,PF 697,PF 698,PF 699,PF 700,PF 701,PF 702,PF 703,PF 704,PF 705,PF 706,PF 707,PF 708,PF 709,PF 710,PF 711,PF 712,PF 713,PF 714,PF 715,PF 716,PF 717,PF 718,PF 719,PF 720,PF 721,PF 722,PF 723,PF 724,PF 725,PF 726,PF 727,PF 728,PF 729,PF 730,PF 731,PF 732,PF 733,PF 734,PF 735
River Rch & RM=Churchill River,Main            ,41243.44
     400     600     800    1000    1200    1400    1600    1800    2000    2200
    2400    2600    2800    3000    3200    3400    3600    3800    4000    4200
    4400    4600    4800    5000    5200    5400    5600    5800    6000    6200
    6400    6600    6800    7000    7200     400     600     800    1000    1200
    1400    1600    1800    2000    2200    2400    2600    2800    3000    3200
    3400    3600    3800    4000    4200    4400    4600    4800    5000    5200
    5400    5600    5800    6000    6200    6400    6600    6800    7000    7200
     400     600     800    1000    1200    1400    1600    1800    2000    2200
    2400    2600    2800    3000    3200    3400    3600    3800    4000    4200
    4400    4600    4800    5000    5200    5400    5600    5800    6000    6200
    6400    6600    6800    7000    7200     400     600     800    1000    1200
    1400    1600    1800    2000    2200    2400    2600    2800    3000    3200
    3400    3600    3800    4000    4200    4400    4600    4800    5000    5200
    5400    5600    5800    6000    6200    6400    6600    6800    7000    7200
     400     600     800    1000    1200    1400    1600    1800    2000    2200
    2400    2600    2800    3000    3200    3400    3600    3800    4000    4200
    4400    4600    4800    5000    5200    5400    5600    5800    6000    6200
    6400    6600    6800    7000    7200     400     600     800    1000    1200
    1400    1600    1800    2000    2200    2400    2600    2800    3000    3200
    3400    3600    3800    4000    4200    4400    4600    4800    5000    5200
    5400    5600    5800    6000    6200    6400    6600    6800    7000    7200
     400     600     800    1000    1200    1400    1600    1800    2000    2200
    2400    2600    2800    3000    3200    3400    3600    3800    4000    4200
    4400    4600    4800    5000    5200    5400    5600    5800    6000    6200
    6400    6600    6800    7000    7200     400     600     800    1000    1200
    1400    1600    1800    2000    2200    2400    2600    2800    3000    3200
    3400    3600    3800    4000    4200    4400    4600    4800    5000    5200
    5400    5600    5800    6000    6200    6400    6600    6800    7000    7200
     400     600     800    1000    1200    1400    1600    1800    2000    2200
    2400    2600    2800    3000    3200    3400    3600    3800    4000    4200
    4400    4600    4800    5000    5200    5400    5600    5800    6000    6200
    6400    6600    6800    7000    7200     400     600     800    1000    1200
    1400    1600    1800    2000    2200    2400    2600    2800    3000    3200
    3400    3600    3800    4000    4200    4400    4600    4800    5000    5200
    5400    5600    5800    6000    6200    6400    6600    6800    7000    7200
     400     600     800    1000    1200    1400    1600    1800    2000    2200
    2400    2600    2800    3000    3200    3400    3600    3800    4000    4200
    4400    4600    4800    5000    5200    5400    5600    5800    6000    6200
    6400    6600    6800    7000    7200     400     600     800    1000    1200
    1400    1600    1800    2000    2200    2400    2600    2800    3000    3200
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Boundary for River Rch & Prof#=Churchill River,Main            , 1
Up Type= 0
Dn Type= 1
Dn Known WS=-1
Boundary for River Rch & Prof#=Churchill River,Main            , 2
Up Type= 0
Dn Type= 1
Dn Known WS=-1
Boundary for River Rch & Prof#=Churchill River,Main            , 3
Up Type= 0
Dn Type= 1
Dn Known WS=-1
Boundary for River Rch & Prof#=Churchill River,Main            , 4
Up Type= 0
Dn Type= 1
Dn Known WS=-1
Boundary for River Rch & Prof#=Churchill River,Main            , 5
Up Type= 0
Dn Type= 1
Dn Known WS=-1
Boundary for River Rch & Prof#=Churchill River,Main            , 6
Up Type= 0
Dn Type= 1
Dn Known WS=-1
Boundary for River Rch & Prof#=Churchill River,Main            , 7
Up Type= 0
Dn Type= 1
Dn Known WS=-1
Boundary for River Rch & Prof#=Churchill River,Main            , 8
Up Type= 0
Dn Type= 1
Dn Known WS=-1
Boundary for River Rch & Prof#=Churchill River,Main            , 9
Up Type= 0
Dn Type= 1
Dn Known WS=-1
Boundary for River Rch & Prof#=Churchill River,Main            , 10
Up Type= 0
Dn Type= 1
Dn Known WS=-1
Boundary for River Rch & Prof#=Churchill River,Main            , 11
Up Type= 0
Dn Type= 1
Dn Known WS=-1
Boundary for River Rch & Prof#=Churchill River,Main            , 12
Up Type= 0
Dn Type= 1
Dn Known WS=-1
Boundary for River Rch & Prof#=Churchill River,Main            , 13
Up Type= 0
Dn Type= 1
Dn Known WS=-1
Boundary for River Rch & Prof#=Churchill River,Main            , 14
Up Type= 0
Dn Type= 1
Dn Known WS=-1
Boundary for River Rch & Prof#=Churchill River,Main            , 15
Up Type= 0
Dn Type= 1
Dn Known WS=-1
Boundary for River Rch & Prof#=Churchill River,Main            , 16
Up Type= 0
Dn Type= 1
Dn Known WS=-1
Boundary for River Rch & Prof#=Churchill River,Main            , 17
Up Type= 0
Dn Type= 1
Dn Known WS=-1
Boundary for River Rch & Prof#=Churchill River,Main            , 18
Up Type= 0
Dn Type= 1
Dn Known WS=-1
Boundary for River Rch & Prof#=Churchill River,Main            , 19
Up Type= 0
Dn Type= 1
Dn Known WS=-1
Boundary for River Rch & Prof#=Churchill River,Main            , 20
Up Type= 0
Dn Type= 1
Dn Known WS=-1
Boundary for River Rch & Prof#=Churchill River,Main            , 21
Up Type= 0
Dn Type= 1
Dn Known WS=-1
Boundary for River Rch & Prof#=Churchill River,Main            , 22
Up Type= 0
Dn Type= 1
Dn Known WS=-1
Boundary for River Rch & Prof#=Churchill River,Main            , 23
Up Type= 0
Dn Type= 1
Dn Known WS=-1
Boundary for River Rch & Prof#=Churchill River,Main            , 24
Up Type= 0
Dn Type= 1
Dn Known WS=-1
Boundary for River Rch & Prof#=Churchill River,Main            , 25
Up Type= 0
Dn Type= 1
Dn Known WS=-1
Boundary for River Rch & Prof#=Churchill River,Main            , 26
Up Type= 0
Dn Type= 1
Dn Known WS=-1
Boundary for River Rch & Prof#=Churchill River,Main            , 27
Up Type= 0
Dn Type= 1
Dn Known WS=-1
Boundary for River Rch & Prof#=Churchill River,Main            , 28
Up Type= 0
Dn Type= 1
Dn Known WS=-1
Boundary for River Rch & Prof#=Churchill River,Main            , 29
Up Type= 0
Dn Type= 1
Dn Known WS=-1
Boundary for River Rch & Prof#=Churchill River,Main            , 30
Up Type= 0
Dn Type= 1
Dn Known WS=-1
Boundary for River Rch & Prof#=Churchill River,Main            , 31
Up Type= 0
Dn Type= 1
Dn Known WS=-1
Boundary for River Rch & Prof#=Churchill River,Main            , 32
Up Type= 0
Dn Type= 1
Dn Known WS=-1
Boundary for River Rch & Prof#=Churchill River,Main            , 33
Up Type= 0
Dn Type= 1
Dn Known WS=-1
Boundary for River Rch & Prof#=Churchill River,Main            , 34
Up Type= 0
Dn Type= 1
Dn Known WS=-1
Boundary for River Rch & Prof#=Churchill River,Main            , 35
Up Type= 0
Dn Type= 1
Dn Known WS=-1
Boundary for River Rch & Prof#=Churchill River,Main            , 36
Up Type= 0
Dn Type= 1
Dn Known WS=-0.9
Boundary for River Rch & Prof#=Churchill River,Main            , 37
Up Type= 0
Dn Type= 1
Dn Known WS=-0.9
Boundary for River Rch & Prof#=Churchill River,Main            , 38
Up Type= 0
Dn Type= 1
Dn Known WS=-0.9
Boundary for River Rch & Prof#=Churchill River,Main            , 39
Up Type= 0
Dn Type= 1
Dn Known WS=-0.9
Boundary for River Rch & Prof#=Churchill River,Main            , 40
Up Type= 0
Dn Type= 1
Dn Known WS=-0.9
Boundary for River Rch & Prof#=Churchill River,Main            , 41
Up Type= 0
Dn Type= 1
Dn Known WS=-0.9
Boundary for River Rch & Prof#=Churchill River,Main            , 42
Up Type= 0
Dn Type= 1
Dn Known WS=-0.9
Boundary for River Rch & Prof#=Churchill River,Main            , 43
Up Type= 0
Dn Type= 1
Dn Known WS=-0.9
Boundary for River Rch & Prof#=Churchill River,Main            , 44
Up Type= 0
Dn Type= 1
Dn Known WS=-0.9
Boundary for River Rch & Prof#=Churchill River,Main            , 45
Up Type= 0
Dn Type= 1
Dn Known WS=-0.9
Boundary for River Rch & Prof#=Churchill River,Main            , 46
Up Type= 0
Dn Type= 1
Dn Known WS=-0.9
Boundary for River Rch & Prof#=Churchill River,Main            , 47
Up Type= 0
Dn Type= 1
Dn Known WS=-0.9
Boundary for River Rch & Prof#=Churchill River,Main            , 48
Up Type= 0
Dn Type= 1
Dn Known WS=-0.9
Boundary for River Rch & Prof#=Churchill River,Main            , 49
Up Type= 0
Dn Type= 1
Dn Known WS=-0.9
Boundary for River Rch & Prof#=Churchill River,Main            , 50
Up Type= 0
Dn Type= 1
Dn Known WS=-0.9
Boundary for River Rch & Prof#=Churchill River,Main            , 51
Up Type= 0
Dn Type= 1
Dn Known WS=-0.9
Boundary for River Rch & Prof#=Churchill River,Main            , 52
Up Type= 0
Dn Type= 1
Dn Known WS=-0.9
Boundary for River Rch & Prof#=Churchill River,Main            , 53
Up Type= 0
Dn Type= 1
Dn Known WS=-0.9
Boundary for River Rch & Prof#=Churchill River,Main            , 54
Up Type= 0
Dn Type= 1
Dn Known WS=-0.9
Boundary for River Rch & Prof#=Churchill River,Main            , 55
Up Type= 0
Dn Type= 1
Dn Known WS=-0.9
Boundary for River Rch & Prof#=Churchill River,Main            , 56
Up Type= 0
Dn Type= 1
Dn Known WS=-0.9
Boundary for River Rch & Prof#=Churchill River,Main            , 57
Up Type= 0
Dn Type= 1
Dn Known WS=-0.9
Boundary for River Rch & Prof#=Churchill River,Main            , 58
Up Type= 0
Dn Type= 1
Dn Known WS=-0.9
Boundary for River Rch & Prof#=Churchill River,Main            , 59
Up Type= 0
Dn Type= 1
Dn Known WS=-0.9
Boundary for River Rch & Prof#=Churchill River,Main            , 60
Up Type= 0
Dn Type= 1
Dn Known WS=-0.9
Boundary for River Rch & Prof#=Churchill River,Main            , 61
Up Type= 0
Dn Type= 1
Dn Known WS=-0.9
Boundary for River Rch & Prof#=Churchill River,Main            , 62
Up Type= 0
Dn Type= 1
Dn Known WS=-0.9
Boundary for River Rch & Prof#=Churchill River,Main            , 63
Up Type= 0
Dn Type= 1
Dn Known WS=-0.9
Boundary for River Rch & Prof#=Churchill River,Main            , 64
Up Type= 0
Dn Type= 1
Dn Known WS=-0.9
Boundary for River Rch & Prof#=Churchill River,Main            , 65
Up Type= 0
Dn Type= 1
Dn Known WS=-0.9
Boundary for River Rch & Prof#=Churchill River,Main            , 66
Up Type= 0
Dn Type= 1
Dn Known WS=-0.9
Boundary for River Rch & Prof#=Churchill River,Main            , 67
Up Type= 0
Dn Type= 1
Dn Known WS=-0.9
Boundary for River Rch & Prof#=Churchill River,Main            , 68
Up Type= 0
Dn Type= 1
Dn Known WS=-0.9
Boundary for River Rch & Prof#=Churchill River,Main            , 69
Up Type= 0
Dn Type= 1
Dn Known WS=-0.9
Boundary for River Rch & Prof#=Churchill River,Main            , 70
Up Type= 0
Dn Type= 1
Dn Known WS=-0.9
Boundary for River Rch & Prof#=Churchill River,Main            , 71
Up Type= 0
Dn Type= 1
Dn Known WS=-0.8
Boundary for River Rch & Prof#=Churchill River,Main            , 72
Up Type= 0
Dn Type= 1
Dn Known WS=-0.8
Boundary for River Rch & Prof#=Churchill River,Main            , 73
Up Type= 0
Dn Type= 1
Dn Known WS=-0.8
Boundary for River Rch & Prof#=Churchill River,Main            , 74
Up Type= 0
Dn Type= 1
Dn Known WS=-0.8
Boundary for River Rch & Prof#=Churchill River,Main            , 75
Up Type= 0
Dn Type= 1
Dn Known WS=-0.8
Boundary for River Rch & Prof#=Churchill River,Main            , 76
Up Type= 0
Dn Type= 1
Dn Known WS=-0.8
Boundary for River Rch & Prof#=Churchill River,Main            , 77
Up Type= 0
Dn Type= 1
Dn Known WS=-0.8
Boundary for River Rch & Prof#=Churchill River,Main            , 78
Up Type= 0
Dn Type= 1
Dn Known WS=-0.8
Boundary for River Rch & Prof#=Churchill River,Main            , 79
Up Type= 0
Dn Type= 1
Dn Known WS=-0.8
Boundary for River Rch & Prof#=Churchill River,Main            , 80
Up Type= 0
Dn Type= 1
Dn Known WS=-0.8
Boundary for River Rch & Prof#=Churchill River,Main            , 81
Up Type= 0
Dn Type= 1
Dn Known WS=-0.8
Boundary for River Rch & Prof#=Churchill River,Main            , 82
Up Type= 0
Dn Type= 1
Dn Known WS=-0.8
Boundary for River Rch & Prof#=Churchill River,Main            , 83
Up Type= 0
Dn Type= 1
Dn Known WS=-0.8
Boundary for River Rch & Prof#=Churchill River,Main            , 84
Up Type= 0
Dn Type= 1
Dn Known WS=-0.8
Boundary for River Rch & Prof#=Churchill River,Main            , 85
Up Type= 0
Dn Type= 1
Dn Known WS=-0.8
Boundary for River Rch & Prof#=Churchill River,Main            , 86
Up Type= 0
Dn Type= 1
Dn Known WS=-0.8
Boundary for River Rch & Prof#=Churchill River,Main            , 87
Up Type= 0
Dn Type= 1
Dn Known WS=-0.8
Boundary for River Rch & Prof#=Churchill River,Main            , 88
Up Type= 0
Dn Type= 1
Dn Known WS=-0.8
Boundary for River Rch & Prof#=Churchill River,Main            , 89
Up Type= 0
Dn Type= 1
Dn Known WS=-0.8
Boundary for River Rch & Prof#=Churchill River,Main            , 90
Up Type= 0
Dn Type= 1
Dn Known WS=-0.8
Boundary for River Rch & Prof#=Churchill River,Main            , 91
Up Type= 0
Dn Type= 1
Dn Known WS=-0.8
Boundary for River Rch & Prof#=Churchill River,Main            , 92
Up Type= 0
Dn Type= 1
Dn Known WS=-0.8
Boundary for River Rch & Prof#=Churchill River,Main            , 93
Up Type= 0
Dn Type= 1
Dn Known WS=-0.8
Boundary for River Rch & Prof#=Churchill River,Main            , 94
Up Type= 0
Dn Type= 1
Dn Known WS=-0.8
Boundary for River Rch & Prof#=Churchill River,Main            , 95
Up Type= 0
Dn Type= 1
Dn Known WS=-0.8
Boundary for River Rch & Prof#=Churchill River,Main            , 96
Up Type= 0
Dn Type= 1
Dn Known WS=-0.8
Boundary for River Rch & Prof#=Churchill River,Main            , 97
Up Type= 0
Dn Type= 1
Dn Known WS=-0.8
Boundary for River Rch & Prof#=Churchill River,Main            , 98
Up Type= 0
Dn Type= 1
Dn Known WS=-0.8
Boundary for River Rch & Prof#=Churchill River,Main            , 99
Up Type= 0
Dn Type= 1
Dn Known WS=-0.8
Boundary for River Rch & Prof#=Churchill River,Main            , 100
Up Type= 0
Dn Type= 1
Dn Known WS=-0.8
Boundary for River Rch & Prof#=Churchill River,Main            , 101
Up Type= 0
Dn Type= 1
Dn Known WS=-0.8
Boundary for River Rch & Prof#=Churchill River,Main            , 102
Up Type= 0
Dn Type= 1
Dn Known WS=-0.8
Boundary for River Rch & Prof#=Churchill River,Main            , 103
Up Type= 0
Dn Type= 1
Dn Known WS=-0.8
Boundary for River Rch & Prof#=Churchill River,Main            , 104
Up Type= 0
Dn Type= 1
Dn Known WS=-0.8
Boundary for River Rch & Prof#=Churchill River,Main            , 105
Up Type= 0
Dn Type= 1
Dn Known WS=-0.8
Boundary for River Rch & Prof#=Churchill River,Main            , 106
Up Type= 0
Dn Type= 1
Dn Known WS=-0.7
Boundary for River Rch & Prof#=Churchill River,Main            , 107
Up Type= 0
Dn Type= 1
Dn Known WS=-0.7
Boundary for River Rch & Prof#=Churchill River,Main            , 108
Up Type= 0
Dn Type= 1
Dn Known WS=-0.7
Boundary for River Rch & Prof#=Churchill River,Main            , 109
Up Type= 0
Dn Type= 1
Dn Known WS=-0.7
Boundary for River Rch & Prof#=Churchill River,Main            , 110
Up Type= 0
Dn Type= 1
Dn Known WS=-0.7
Boundary for River Rch & Prof#=Churchill River,Main            , 111
Up Type= 0
Dn Type= 1
Dn Known WS=-0.7
Boundary for River Rch & Prof#=Churchill River,Main            , 112
Up Type= 0
Dn Type= 1
Dn Known WS=-0.7
Boundary for River Rch & Prof#=Churchill River,Main            , 113
Up Type= 0
Dn Type= 1
Dn Known WS=-0.7
Boundary for River Rch & Prof#=Churchill River,Main            , 114
Up Type= 0
Dn Type= 1
Dn Known WS=-0.7
Boundary for River Rch & Prof#=Churchill River,Main            , 115
Up Type= 0
Dn Type= 1
Dn Known WS=-0.7
Boundary for River Rch & Prof#=Churchill River,Main            , 116
Up Type= 0
Dn Type= 1
Dn Known WS=-0.7
Boundary for River Rch & Prof#=Churchill River,Main            , 117
Up Type= 0
Dn Type= 1
Dn Known WS=-0.7
Boundary for River Rch & Prof#=Churchill River,Main            , 118
Up Type= 0
Dn Type= 1
Dn Known WS=-0.7
Boundary for River Rch & Prof#=Churchill River,Main            , 119
Up Type= 0
Dn Type= 1
Dn Known WS=-0.7
Boundary for River Rch & Prof#=Churchill River,Main            , 120
Up Type= 0
Dn Type= 1
Dn Known WS=-0.7
Boundary for River Rch & Prof#=Churchill River,Main            , 121
Up Type= 0
Dn Type= 1
Dn Known WS=-0.7
Boundary for River Rch & Prof#=Churchill River,Main            , 122
Up Type= 0
Dn Type= 1
Dn Known WS=-0.7
Boundary for River Rch & Prof#=Churchill River,Main            , 123
Up Type= 0
Dn Type= 1
Dn Known WS=-0.7
Boundary for River Rch & Prof#=Churchill River,Main            , 124
Up Type= 0
Dn Type= 1
Dn Known WS=-0.7
Boundary for River Rch & Prof#=Churchill River,Main            , 125
Up Type= 0
Dn Type= 1
Dn Known WS=-0.7
Boundary for River Rch & Prof#=Churchill River,Main            , 126
Up Type= 0
Dn Type= 1
Dn Known WS=-0.7
Boundary for River Rch & Prof#=Churchill River,Main            , 127
Up Type= 0
Dn Type= 1
Dn Known WS=-0.7
Boundary for River Rch & Prof#=Churchill River,Main            , 128
Up Type= 0
Dn Type= 1
Dn Known WS=-0.7
Boundary for River Rch & Prof#=Churchill River,Main            , 129
Up Type= 0
Dn Type= 1
Dn Known WS=-0.7
Boundary for River Rch & Prof#=Churchill River,Main            , 130
Up Type= 0
Dn Type= 1
Dn Known WS=-0.7
Boundary for River Rch & Prof#=Churchill River,Main            , 131
Up Type= 0
Dn Type= 1
Dn Known WS=-0.7
Boundary for River Rch & Prof#=Churchill River,Main            , 132
Up Type= 0
Dn Type= 1
Dn Known WS=-0.7
Boundary for River Rch & Prof#=Churchill River,Main            , 133
Up Type= 0
Dn Type= 1
Dn Known WS=-0.7
Boundary for River Rch & Prof#=Churchill River,Main            , 134
Up Type= 0
Dn Type= 1
Dn Known WS=-0.7
Boundary for River Rch & Prof#=Churchill River,Main            , 135
Up Type= 0
Dn Type= 1
Dn Known WS=-0.7
Boundary for River Rch & Prof#=Churchill River,Main            , 136
Up Type= 0
Dn Type= 1
Dn Known WS=-0.7
Boundary for River Rch & Prof#=Churchill River,Main            , 137
Up Type= 0
Dn Type= 1
Dn Known WS=-0.7
Boundary for River Rch & Prof#=Churchill River,Main            , 138
Up Type= 0
Dn Type= 1
Dn Known WS=-0.7
Boundary for River Rch & Prof#=Churchill River,Main            , 139
Up Type= 0
Dn Type= 1
Dn Known WS=-0.7
Boundary for River Rch & Prof#=Churchill River,Main            , 140
Up Type= 0
Dn Type= 1
Dn Known WS=-0.7
Boundary for River Rch & Prof#=Churchill River,Main            , 141
Up Type= 0
Dn Type= 1
Dn Known WS=-0.6
Boundary for River Rch & Prof#=Churchill River,Main            , 142
Up Type= 0
Dn Type= 1
Dn Known WS=-0.6
Boundary for River Rch & Prof#=Churchill River,Main            , 143
Up Type= 0
Dn Type= 1
Dn Known WS=-0.6
Boundary for River Rch & Prof#=Churchill River,Main            , 144
Up Type= 0
Dn Type= 1
Dn Known WS=-0.6
Boundary for River Rch & Prof#=Churchill River,Main            , 145
Up Type= 0
Dn Type= 1
Dn Known WS=-0.6
Boundary for River Rch & Prof#=Churchill River,Main            , 146
Up Type= 0
Dn Type= 1
Dn Known WS=-0.6
Boundary for River Rch & Prof#=Churchill River,Main            , 147
Up Type= 0
Dn Type= 1
Dn Known WS=-0.6
Boundary for River Rch & Prof#=Churchill River,Main            , 148
Up Type= 0
Dn Type= 1
Dn Known WS=-0.6
Boundary for River Rch & Prof#=Churchill River,Main            , 149
Up Type= 0
Dn Type= 1
Dn Known WS=-0.6
Boundary for River Rch & Prof#=Churchill River,Main            , 150
Up Type= 0
Dn Type= 1
Dn Known WS=-0.6
Boundary for River Rch & Prof#=Churchill River,Main            , 151
Up Type= 0
Dn Type= 1
Dn Known WS=-0.6
Boundary for River Rch & Prof#=Churchill River,Main            , 152
Up Type= 0
Dn Type= 1
Dn Known WS=-0.6
Boundary for River Rch & Prof#=Churchill River,Main            , 153
Up Type= 0
Dn Type= 1
Dn Known WS=-0.6
Boundary for River Rch & Prof#=Churchill River,Main            , 154
Up Type= 0
Dn Type= 1
Dn Known WS=-0.6
Boundary for River Rch & Prof#=Churchill River,Main            , 155
Up Type= 0
Dn Type= 1
Dn Known WS=-0.6
Boundary for River Rch & Prof#=Churchill River,Main            , 156
Up Type= 0
Dn Type= 1
Dn Known WS=-0.6
Boundary for River Rch & Prof#=Churchill River,Main            , 157
Up Type= 0
Dn Type= 1
Dn Known WS=-0.6
Boundary for River Rch & Prof#=Churchill River,Main            , 158
Up Type= 0
Dn Type= 1
Dn Known WS=-0.6
Boundary for River Rch & Prof#=Churchill River,Main            , 159
Up Type= 0
Dn Type= 1
Dn Known WS=-0.6
Boundary for River Rch & Prof#=Churchill River,Main            , 160
Up Type= 0
Dn Type= 1
Dn Known WS=-0.6
Boundary for River Rch & Prof#=Churchill River,Main            , 161
Up Type= 0
Dn Type= 1
Dn Known WS=-0.6
Boundary for River Rch & Prof#=Churchill River,Main            , 162
Up Type= 0
Dn Type= 1
Dn Known WS=-0.6
Boundary for River Rch & Prof#=Churchill River,Main            , 163
Up Type= 0
Dn Type= 1
Dn Known WS=-0.6
Boundary for River Rch & Prof#=Churchill River,Main            , 164
Up Type= 0
Dn Type= 1
Dn Known WS=-0.6
Boundary for River Rch & Prof#=Churchill River,Main            , 165
Up Type= 0
Dn Type= 1
Dn Known WS=-0.6
Boundary for River Rch & Prof#=Churchill River,Main            , 166
Up Type= 0
Dn Type= 1
Dn Known WS=-0.6
Boundary for River Rch & Prof#=Churchill River,Main            , 167
Up Type= 0
Dn Type= 1
Dn Known WS=-0.6
Boundary for River Rch & Prof#=Churchill River,Main            , 168
Up Type= 0
Dn Type= 1
Dn Known WS=-0.6
Boundary for River Rch & Prof#=Churchill River,Main            , 169
Up Type= 0
Dn Type= 1
Dn Known WS=-0.6
Boundary for River Rch & Prof#=Churchill River,Main            , 170
Up Type= 0
Dn Type= 1
Dn Known WS=-0.6
Boundary for River Rch & Prof#=Churchill River,Main            , 171
Up Type= 0
Dn Type= 1
Dn Known WS=-0.6
Boundary for River Rch & Prof#=Churchill River,Main            , 172
Up Type= 0
Dn Type= 1
Dn Known WS=-0.6
Boundary for River Rch & Prof#=Churchill River,Main            , 173
Up Type= 0
Dn Type= 1
Dn Known WS=-0.6
Boundary for River Rch & Prof#=Churchill River,Main            , 174
Up Type= 0
Dn Type= 1
Dn Known WS=-0.6
Boundary for River Rch & Prof#=Churchill River,Main            , 175
Up Type= 0
Dn Type= 1
Dn Known WS=-0.6
Boundary for River Rch & Prof#=Churchill River,Main            , 176
Up Type= 0
Dn Type= 1
Dn Known WS=-0.5
Boundary for River Rch & Prof#=Churchill River,Main            , 177
Up Type= 0
Dn Type= 1
Dn Known WS=-0.5
Boundary for River Rch & Prof#=Churchill River,Main            , 178
Up Type= 0
Dn Type= 1
Dn Known WS=-0.5
Boundary for River Rch & Prof#=Churchill River,Main            , 179
Up Type= 0
Dn Type= 1
Dn Known WS=-0.5
Boundary for River Rch & Prof#=Churchill River,Main            , 180
Up Type= 0
Dn Type= 1
Dn Known WS=-0.5
Boundary for River Rch & Prof#=Churchill River,Main            , 181
Up Type= 0
Dn Type= 1
Dn Known WS=-0.5
Boundary for River Rch & Prof#=Churchill River,Main            , 182
Up Type= 0
Dn Type= 1
Dn Known WS=-0.5
Boundary for River Rch & Prof#=Churchill River,Main            , 183
Up Type= 0
Dn Type= 1
Dn Known WS=-0.5
Boundary for River Rch & Prof#=Churchill River,Main            , 184
Up Type= 0
Dn Type= 1
Dn Known WS=-0.5
Boundary for River Rch & Prof#=Churchill River,Main            , 185
Up Type= 0
Dn Type= 1
Dn Known WS=-0.5
Boundary for River Rch & Prof#=Churchill River,Main            , 186
Up Type= 0
Dn Type= 1
Dn Known WS=-0.5
Boundary for River Rch & Prof#=Churchill River,Main            , 187
Up Type= 0
Dn Type= 1
Dn Known WS=-0.5
Boundary for River Rch & Prof#=Churchill River,Main            , 188
Up Type= 0
Dn Type= 1
Dn Known WS=-0.5
Boundary for River Rch & Prof#=Churchill River,Main            , 189
Up Type= 0
Dn Type= 1
Dn Known WS=-0.5
Boundary for River Rch & Prof#=Churchill River,Main            , 190
Up Type= 0
Dn Type= 1
Dn Known WS=-0.5
Boundary for River Rch & Prof#=Churchill River,Main            , 191
Up Type= 0
Dn Type= 1
Dn Known WS=-0.5
Boundary for River Rch & Prof#=Churchill River,Main            , 192
Up Type= 0
Dn Type= 1
Dn Known WS=-0.5
Boundary for River Rch & Prof#=Churchill River,Main            , 193
Up Type= 0
Dn Type= 1
Dn Known WS=-0.5
Boundary for River Rch & Prof#=Churchill River,Main            , 194
Up Type= 0
Dn Type= 1
Dn Known WS=-0.5
Boundary for River Rch & Prof#=Churchill River,Main            , 195
Up Type= 0
Dn Type= 1
Dn Known WS=-0.5
Boundary for River Rch & Prof#=Churchill River,Main            , 196
Up Type= 0
Dn Type= 1
Dn Known WS=-0.5
Boundary for River Rch & Prof#=Churchill River,Main            , 197
Up Type= 0
Dn Type= 1
Dn Known WS=-0.5
Boundary for River Rch & Prof#=Churchill River,Main            , 198
Up Type= 0
Dn Type= 1
Dn Known WS=-0.5
Boundary for River Rch & Prof#=Churchill River,Main            , 199
Up Type= 0
Dn Type= 1
Dn Known WS=-0.5
Boundary for River Rch & Prof#=Churchill River,Main            , 200
Up Type= 0
Dn Type= 1
Dn Known WS=-0.5
Boundary for River Rch & Prof#=Churchill River,Main            , 201
Up Type= 0
Dn Type= 1
Dn Known WS=-0.5
Boundary for River Rch & Prof#=Churchill River,Main            , 202
Up Type= 0
Dn Type= 1
Dn Known WS=-0.5
Boundary for River Rch & Prof#=Churchill River,Main            , 203
Up Type= 0
Dn Type= 1
Dn Known WS=-0.5
Boundary for River Rch & Prof#=Churchill River,Main            , 204
Up Type= 0
Dn Type= 1
Dn Known WS=-0.5
Boundary for River Rch & Prof#=Churchill River,Main            , 205
Up Type= 0
Dn Type= 1
Dn Known WS=-0.5
Boundary for River Rch & Prof#=Churchill River,Main            , 206
Up Type= 0
Dn Type= 1
Dn Known WS=-0.5
Boundary for River Rch & Prof#=Churchill River,Main            , 207
Up Type= 0
Dn Type= 1
Dn Known WS=-0.5
Boundary for River Rch & Prof#=Churchill River,Main            , 208
Up Type= 0
Dn Type= 1
Dn Known WS=-0.5
Boundary for River Rch & Prof#=Churchill River,Main            , 209
Up Type= 0
Dn Type= 1
Dn Known WS=-0.5
Boundary for River Rch & Prof#=Churchill River,Main            , 210
Up Type= 0
Dn Type= 1
Dn Known WS=-0.5
Boundary for River Rch & Prof#=Churchill River,Main            , 211
Up Type= 0
Dn Type= 1
Dn Known WS=-0.4
Boundary for River Rch & Prof#=Churchill River,Main            , 212
Up Type= 0
Dn Type= 1
Dn Known WS=-0.4
Boundary for River Rch & Prof#=Churchill River,Main            , 213
Up Type= 0
Dn Type= 1
Dn Known WS=-0.4
Boundary for River Rch & Prof#=Churchill River,Main            , 214
Up Type= 0
Dn Type= 1
Dn Known WS=-0.4
Boundary for River Rch & Prof#=Churchill River,Main            , 215
Up Type= 0
Dn Type= 1
Dn Known WS=-0.4
Boundary for River Rch & Prof#=Churchill River,Main            , 216
Up Type= 0
Dn Type= 1
Dn Known WS=-0.4
Boundary for River Rch & Prof#=Churchill River,Main            , 217
Up Type= 0
Dn Type= 1
Dn Known WS=-0.4
Boundary for River Rch & Prof#=Churchill River,Main            , 218
Up Type= 0
Dn Type= 1
Dn Known WS=-0.4
Boundary for River Rch & Prof#=Churchill River,Main            , 219
Up Type= 0
Dn Type= 1
Dn Known WS=-0.4
Boundary for River Rch & Prof#=Churchill River,Main            , 220
Up Type= 0
Dn Type= 1
Dn Known WS=-0.4
Boundary for River Rch & Prof#=Churchill River,Main            , 221
Up Type= 0
Dn Type= 1
Dn Known WS=-0.4
Boundary for River Rch & Prof#=Churchill River,Main            , 222
Up Type= 0
Dn Type= 1
Dn Known WS=-0.4
Boundary for River Rch & Prof#=Churchill River,Main            , 223
Up Type= 0
Dn Type= 1
Dn Known WS=-0.4
Boundary for River Rch & Prof#=Churchill River,Main            , 224
Up Type= 0
Dn Type= 1
Dn Known WS=-0.4
Boundary for River Rch & Prof#=Churchill River,Main            , 225
Up Type= 0
Dn Type= 1
Dn Known WS=-0.4
Boundary for River Rch & Prof#=Churchill River,Main            , 226
Up Type= 0
Dn Type= 1
Dn Known WS=-0.4
Boundary for River Rch & Prof#=Churchill River,Main            , 227
Up Type= 0
Dn Type= 1
Dn Known WS=-0.4
Boundary for River Rch & Prof#=Churchill River,Main            , 228
Up Type= 0
Dn Type= 1
Dn Known WS=-0.4
Boundary for River Rch & Prof#=Churchill River,Main            , 229
Up Type= 0
Dn Type= 1
Dn Known WS=-0.4
Boundary for River Rch & Prof#=Churchill River,Main            , 230
Up Type= 0
Dn Type= 1
Dn Known WS=-0.4
Boundary for River Rch & Prof#=Churchill River,Main            , 231
Up Type= 0
Dn Type= 1
Dn Known WS=-0.4
Boundary for River Rch & Prof#=Churchill River,Main            , 232
Up Type= 0
Dn Type= 1
Dn Known WS=-0.4
Boundary for River Rch & Prof#=Churchill River,Main            , 233
Up Type= 0
Dn Type= 1
Dn Known WS=-0.4
Boundary for River Rch & Prof#=Churchill River,Main            , 234
Up Type= 0
Dn Type= 1
Dn Known WS=-0.4
Boundary for River Rch & Prof#=Churchill River,Main            , 235
Up Type= 0
Dn Type= 1
Dn Known WS=-0.4
Boundary for River Rch & Prof#=Churchill River,Main            , 236
Up Type= 0
Dn Type= 1
Dn Known WS=-0.4
Boundary for River Rch & Prof#=Churchill River,Main            , 237
Up Type= 0
Dn Type= 1
Dn Known WS=-0.4
Boundary for River Rch & Prof#=Churchill River,Main            , 238
Up Type= 0
Dn Type= 1
Dn Known WS=-0.4
Boundary for River Rch & Prof#=Churchill River,Main            , 239
Up Type= 0
Dn Type= 1
Dn Known WS=-0.4
Boundary for River Rch & Prof#=Churchill River,Main            , 240
Up Type= 0
Dn Type= 1
Dn Known WS=-0.4
Boundary for River Rch & Prof#=Churchill River,Main            , 241
Up Type= 0
Dn Type= 1
Dn Known WS=-0.4
Boundary for River Rch & Prof#=Churchill River,Main            , 242
Up Type= 0
Dn Type= 1
Dn Known WS=-0.4
Boundary for River Rch & Prof#=Churchill River,Main            , 243
Up Type= 0
Dn Type= 1
Dn Known WS=-0.4
Boundary for River Rch & Prof#=Churchill River,Main            , 244
Up Type= 0
Dn Type= 1
Dn Known WS=-0.4
Boundary for River Rch & Prof#=Churchill River,Main            , 245
Up Type= 0
Dn Type= 1
Dn Known WS=-0.4
Boundary for River Rch & Prof#=Churchill River,Main            , 246
Up Type= 0
Dn Type= 1
Dn Known WS=-0.3
Boundary for River Rch & Prof#=Churchill River,Main            , 247
Up Type= 0
Dn Type= 1
Dn Known WS=-0.3
Boundary for River Rch & Prof#=Churchill River,Main            , 248
Up Type= 0
Dn Type= 1
Dn Known WS=-0.3
Boundary for River Rch & Prof#=Churchill River,Main            , 249
Up Type= 0
Dn Type= 1
Dn Known WS=-0.3
Boundary for River Rch & Prof#=Churchill River,Main            , 250
Up Type= 0
Dn Type= 1
Dn Known WS=-0.3
Boundary for River Rch & Prof#=Churchill River,Main            , 251
Up Type= 0
Dn Type= 1
Dn Known WS=-0.3
Boundary for River Rch & Prof#=Churchill River,Main            , 252
Up Type= 0
Dn Type= 1
Dn Known WS=-0.3
Boundary for River Rch & Prof#=Churchill River,Main            , 253
Up Type= 0
Dn Type= 1
Dn Known WS=-0.3
Boundary for River Rch & Prof#=Churchill River,Main            , 254
Up Type= 0
Dn Type= 1
Dn Known WS=-0.3
Boundary for River Rch & Prof#=Churchill River,Main            , 255
Up Type= 0
Dn Type= 1
Dn Known WS=-0.3
Boundary for River Rch & Prof#=Churchill River,Main            , 256
Up Type= 0
Dn Type= 1
Dn Known WS=-0.3
Boundary for River Rch & Prof#=Churchill River,Main            , 257
Up Type= 0
Dn Type= 1
Dn Known WS=-0.3
Boundary for River Rch & Prof#=Churchill River,Main            , 258
Up Type= 0
Dn Type= 1
Dn Known WS=-0.3
Boundary for River Rch & Prof#=Churchill River,Main            , 259
Up Type= 0
Dn Type= 1
Dn Known WS=-0.3
Boundary for River Rch & Prof#=Churchill River,Main            , 260
Up Type= 0
Dn Type= 1
Dn Known WS=-0.3
Boundary for River Rch & Prof#=Churchill River,Main            , 261
Up Type= 0
Dn Type= 1
Dn Known WS=-0.3
Boundary for River Rch & Prof#=Churchill River,Main            , 262
Up Type= 0
Dn Type= 1
Dn Known WS=-0.3
Boundary for River Rch & Prof#=Churchill River,Main            , 263
Up Type= 0
Dn Type= 1
Dn Known WS=-0.3
Boundary for River Rch & Prof#=Churchill River,Main            , 264
Up Type= 0
Dn Type= 1
Dn Known WS=-0.3
Boundary for River Rch & Prof#=Churchill River,Main            , 265
Up Type= 0
Dn Type= 1
Dn Known WS=-0.3
Boundary for River Rch & Prof#=Churchill River,Main            , 266
Up Type= 0
Dn Type= 1
Dn Known WS=-0.3
Boundary for River Rch & Prof#=Churchill River,Main            , 267
Up Type= 0
Dn Type= 1
Dn Known WS=-0.3
Boundary for River Rch & Prof#=Churchill River,Main            , 268
Up Type= 0
Dn Type= 1
Dn Known WS=-0.3
Boundary for River Rch & Prof#=Churchill River,Main            , 269
Up Type= 0
Dn Type= 1
Dn Known WS=-0.3
Boundary for River Rch & Prof#=Churchill River,Main            , 270
Up Type= 0
Dn Type= 1
Dn Known WS=-0.3
Boundary for River Rch & Prof#=Churchill River,Main            , 271
Up Type= 0
Dn Type= 1
Dn Known WS=-0.3
Boundary for River Rch & Prof#=Churchill River,Main            , 272
Up Type= 0
Dn Type= 1
Dn Known WS=-0.3
Boundary for River Rch & Prof#=Churchill River,Main            , 273
Up Type= 0
Dn Type= 1
Dn Known WS=-0.3
Boundary for River Rch & Prof#=Churchill River,Main            , 274
Up Type= 0
Dn Type= 1
Dn Known WS=-0.3
Boundary for River Rch & Prof#=Churchill River,Main            , 275
Up Type= 0
Dn Type= 1
Dn Known WS=-0.3
Boundary for River Rch & Prof#=Churchill River,Main            , 276
Up Type= 0
Dn Type= 1
Dn Known WS=-0.3
Boundary for River Rch & Prof#=Churchill River,Main            , 277
Up Type= 0
Dn Type= 1
Dn Known WS=-0.3
Boundary for River Rch & Prof#=Churchill River,Main            , 278
Up Type= 0
Dn Type= 1
Dn Known WS=-0.3
Boundary for River Rch & Prof#=Churchill River,Main            , 279
Up Type= 0
Dn Type= 1
Dn Known WS=-0.3
Boundary for River Rch & Prof#=Churchill River,Main            , 280
Up Type= 0
Dn Type= 1
Dn Known WS=-0.3
Boundary for River Rch & Prof#=Churchill River,Main            , 281
Up Type= 0
Dn Type= 1
Dn Known WS=-0.2
Boundary for River Rch & Prof#=Churchill River,Main            , 282
Up Type= 0
Dn Type= 1
Dn Known WS=-0.2
Boundary for River Rch & Prof#=Churchill River,Main            , 283
Up Type= 0
Dn Type= 1
Dn Known WS=-0.2
Boundary for River Rch & Prof#=Churchill River,Main            , 284
Up Type= 0
Dn Type= 1
Dn Known WS=-0.2
Boundary for River Rch & Prof#=Churchill River,Main            , 285
Up Type= 0
Dn Type= 1
Dn Known WS=-0.2
Boundary for River Rch & Prof#=Churchill River,Main            , 286
Up Type= 0
Dn Type= 1
Dn Known WS=-0.2
Boundary for River Rch & Prof#=Churchill River,Main            , 287
Up Type= 0
Dn Type= 1
Dn Known WS=-0.2
Boundary for River Rch & Prof#=Churchill River,Main            , 288
Up Type= 0
Dn Type= 1
Dn Known WS=-0.2
Boundary for River Rch & Prof#=Churchill River,Main            , 289
Up Type= 0
Dn Type= 1
Dn Known WS=-0.2
Boundary for River Rch & Prof#=Churchill River,Main            , 290
Up Type= 0
Dn Type= 1
Dn Known WS=-0.2
Boundary for River Rch & Prof#=Churchill River,Main            , 291
Up Type= 0
Dn Type= 1
Dn Known WS=-0.2
Boundary for River Rch & Prof#=Churchill River,Main            , 292
Up Type= 0
Dn Type= 1
Dn Known WS=-0.2
Boundary for River Rch & Prof#=Churchill River,Main            , 293
Up Type= 0
Dn Type= 1
Dn Known WS=-0.2
Boundary for River Rch & Prof#=Churchill River,Main            , 294
Up Type= 0
Dn Type= 1
Dn Known WS=-0.2
Boundary for River Rch & Prof#=Churchill River,Main            , 295
Up Type= 0
Dn Type= 1
Dn Known WS=-0.2
Boundary for River Rch & Prof#=Churchill River,Main            , 296
Up Type= 0
Dn Type= 1
Dn Known WS=-0.2
Boundary for River Rch & Prof#=Churchill River,Main            , 297
Up Type= 0
Dn Type= 1
Dn Known WS=-0.2
Boundary for River Rch & Prof#=Churchill River,Main            , 298
Up Type= 0
Dn Type= 1
Dn Known WS=-0.2
Boundary for River Rch & Prof#=Churchill River,Main            , 299
Up Type= 0
Dn Type= 1
Dn Known WS=-0.2
Boundary for River Rch & Prof#=Churchill River,Main            , 300
Up Type= 0
Dn Type= 1
Dn Known WS=-0.2
Boundary for River Rch & Prof#=Churchill River,Main            , 301
Up Type= 0
Dn Type= 1
Dn Known WS=-0.2
Boundary for River Rch & Prof#=Churchill River,Main            , 302
Up Type= 0
Dn Type= 1
Dn Known WS=-0.2
Boundary for River Rch & Prof#=Churchill River,Main            , 303
Up Type= 0
Dn Type= 1
Dn Known WS=-0.2
Boundary for River Rch & Prof#=Churchill River,Main            , 304
Up Type= 0
Dn Type= 1
Dn Known WS=-0.2
Boundary for River Rch & Prof#=Churchill River,Main            , 305
Up Type= 0
Dn Type= 1
Dn Known WS=-0.2
Boundary for River Rch & Prof#=Churchill River,Main            , 306
Up Type= 0
Dn Type= 1
Dn Known WS=-0.2
Boundary for River Rch & Prof#=Churchill River,Main            , 307
Up Type= 0
Dn Type= 1
Dn Known WS=-0.2
Boundary for River Rch & Prof#=Churchill River,Main            , 308
Up Type= 0
Dn Type= 1
Dn Known WS=-0.2
Boundary for River Rch & Prof#=Churchill River,Main            , 309
Up Type= 0
Dn Type= 1
Dn Known WS=-0.2
Boundary for River Rch & Prof#=Churchill River,Main            , 310
Up Type= 0
Dn Type= 1
Dn Known WS=-0.2
Boundary for River Rch & Prof#=Churchill River,Main            , 311
Up Type= 0
Dn Type= 1
Dn Known WS=-0.2
Boundary for River Rch & Prof#=Churchill River,Main            , 312
Up Type= 0
Dn Type= 1
Dn Known WS=-0.2
Boundary for River Rch & Prof#=Churchill River,Main            , 313
Up Type= 0
Dn Type= 1
Dn Known WS=-0.2
Boundary for River Rch & Prof#=Churchill River,Main            , 314
Up Type= 0
Dn Type= 1
Dn Known WS=-0.2
Boundary for River Rch & Prof#=Churchill River,Main            , 315
Up Type= 0
Dn Type= 1
Dn Known WS=-0.2
Boundary for River Rch & Prof#=Churchill River,Main            , 316
Up Type= 0
Dn Type= 1
Dn Known WS=-0.1
Boundary for River Rch & Prof#=Churchill River,Main            , 317
Up Type= 0
Dn Type= 1
Dn Known WS=-0.1
Boundary for River Rch & Prof#=Churchill River,Main            , 318
Up Type= 0
Dn Type= 1
Dn Known WS=-0.1
Boundary for River Rch & Prof#=Churchill River,Main            , 319
Up Type= 0
Dn Type= 1
Dn Known WS=-0.1
Boundary for River Rch & Prof#=Churchill River,Main            , 320
Up Type= 0
Dn Type= 1
Dn Known WS=-0.1
Boundary for River Rch & Prof#=Churchill River,Main            , 321
Up Type= 0
Dn Type= 1
Dn Known WS=-0.1
Boundary for River Rch & Prof#=Churchill River,Main            , 322
Up Type= 0
Dn Type= 1
Dn Known WS=-0.1
Boundary for River Rch & Prof#=Churchill River,Main            , 323
Up Type= 0
Dn Type= 1
Dn Known WS=-0.1
Boundary for River Rch & Prof#=Churchill River,Main            , 324
Up Type= 0
Dn Type= 1
Dn Known WS=-0.1
Boundary for River Rch & Prof#=Churchill River,Main            , 325
Up Type= 0
Dn Type= 1
Dn Known WS=-0.1
Boundary for River Rch & Prof#=Churchill River,Main            , 326
Up Type= 0
Dn Type= 1
Dn Known WS=-0.1
Boundary for River Rch & Prof#=Churchill River,Main            , 327
Up Type= 0
Dn Type= 1
Dn Known WS=-0.1
Boundary for River Rch & Prof#=Churchill River,Main            , 328
Up Type= 0
Dn Type= 1
Dn Known WS=-0.1
Boundary for River Rch & Prof#=Churchill River,Main            , 329
Up Type= 0
Dn Type= 1
Dn Known WS=-0.1
Boundary for River Rch & Prof#=Churchill River,Main            , 330
Up Type= 0
Dn Type= 1
Dn Known WS=-0.1
Boundary for River Rch & Prof#=Churchill River,Main            , 331
Up Type= 0
Dn Type= 1
Dn Known WS=-0.1
Boundary for River Rch & Prof#=Churchill River,Main            , 332
Up Type= 0
Dn Type= 1
Dn Known WS=-0.1
Boundary for River Rch & Prof#=Churchill River,Main            , 333
Up Type= 0
Dn Type= 1
Dn Known WS=-0.1
Boundary for River Rch & Prof#=Churchill River,Main            , 334
Up Type= 0
Dn Type= 1
Dn Known WS=-0.1
Boundary for River Rch & Prof#=Churchill River,Main            , 335
Up Type= 0
Dn Type= 1
Dn Known WS=-0.1
Boundary for River Rch & Prof#=Churchill River,Main            , 336
Up Type= 0
Dn Type= 1
Dn Known WS=-0.1
Boundary for River Rch & Prof#=Churchill River,Main            , 337
Up Type= 0
Dn Type= 1
Dn Known WS=-0.1
Boundary for River Rch & Prof#=Churchill River,Main            , 338
Up Type= 0
Dn Type= 1
Dn Known WS=-0.1
Boundary for River Rch & Prof#=Churchill River,Main            , 339
Up Type= 0
Dn Type= 1
Dn Known WS=-0.1
Boundary for River Rch & Prof#=Churchill River,Main            , 340
Up Type= 0
Dn Type= 1
Dn Known WS=-0.1
Boundary for River Rch & Prof#=Churchill River,Main            , 341
Up Type= 0
Dn Type= 1
Dn Known WS=-0.1
Boundary for River Rch & Prof#=Churchill River,Main            , 342
Up Type= 0
Dn Type= 1
Dn Known WS=-0.1
Boundary for River Rch & Prof#=Churchill River,Main            , 343
Up Type= 0
Dn Type= 1
Dn Known WS=-0.1
Boundary for River Rch & Prof#=Churchill River,Main            , 344
Up Type= 0
Dn Type= 1
Dn Known WS=-0.1
Boundary for River Rch & Prof#=Churchill River,Main            , 345
Up Type= 0
Dn Type= 1
Dn Known WS=-0.1
Boundary for River Rch & Prof#=Churchill River,Main            , 346
Up Type= 0
Dn Type= 1
Dn Known WS=-0.1
Boundary for River Rch & Prof#=Churchill River,Main            , 347
Up Type= 0
Dn Type= 1
Dn Known WS=-0.1
Boundary for River Rch & Prof#=Churchill River,Main            , 348
Up Type= 0
Dn Type= 1
Dn Known WS=-0.1
Boundary for River Rch & Prof#=Churchill River,Main            , 349
Up Type= 0
Dn Type= 1
Dn Known WS=-0.1
Boundary for River Rch & Prof#=Churchill River,Main            , 350
Up Type= 0
Dn Type= 1
Dn Known WS=-0.1
Boundary for River Rch & Prof#=Churchill River,Main            , 351
Up Type= 0
Dn Type= 1
Dn Known WS=-1.38778E-16
Boundary for River Rch & Prof#=Churchill River,Main            , 352
Up Type= 0
Dn Type= 1
Dn Known WS=-1.38778E-16
Boundary for River Rch & Prof#=Churchill River,Main            , 353
Up Type= 0
Dn Type= 1
Dn Known WS=-1.38778E-16
Boundary for River Rch & Prof#=Churchill River,Main            , 354
Up Type= 0
Dn Type= 1
Dn Known WS=-1.38778E-16
Boundary for River Rch & Prof#=Churchill River,Main            , 355
Up Type= 0
Dn Type= 1
Dn Known WS=-1.38778E-16
Boundary for River Rch & Prof#=Churchill River,Main            , 356
Up Type= 0
Dn Type= 1
Dn Known WS=-1.38778E-16
Boundary for River Rch & Prof#=Churchill River,Main            , 357
Up Type= 0
Dn Type= 1
Dn Known WS=-1.38778E-16
Boundary for River Rch & Prof#=Churchill River,Main            , 358
Up Type= 0
Dn Type= 1
Dn Known WS=-1.38778E-16
Boundary for River Rch & Prof#=Churchill River,Main            , 359
Up Type= 0
Dn Type= 1
Dn Known WS=-1.38778E-16
Boundary for River Rch & Prof#=Churchill River,Main            , 360
Up Type= 0
Dn Type= 1
Dn Known WS=-1.38778E-16
Boundary for River Rch & Prof#=Churchill River,Main            , 361
Up Type= 0
Dn Type= 1
Dn Known WS=-1.38778E-16
Boundary for River Rch & Prof#=Churchill River,Main            , 362
Up Type= 0
Dn Type= 1
Dn Known WS=-1.38778E-16
Boundary for River Rch & Prof#=Churchill River,Main            , 363
Up Type= 0
Dn Type= 1
Dn Known WS=-1.38778E-16
Boundary for River Rch & Prof#=Churchill River,Main            , 364
Up Type= 0
Dn Type= 1
Dn Known WS=-1.38778E-16
Boundary for River Rch & Prof#=Churchill River,Main            , 365
Up Type= 0
Dn Type= 1
Dn Known WS=-1.38778E-16
Boundary for River Rch & Prof#=Churchill River,Main            , 366
Up Type= 0
Dn Type= 1
Dn Known WS=-1.38778E-16
Boundary for River Rch & Prof#=Churchill River,Main            , 367
Up Type= 0
Dn Type= 1
Dn Known WS=-1.38778E-16
Boundary for River Rch & Prof#=Churchill River,Main            , 368
Up Type= 0
Dn Type= 1
Dn Known WS=-1.38778E-16
Boundary for River Rch & Prof#=Churchill River,Main            , 369
Up Type= 0
Dn Type= 1
Dn Known WS=-1.38778E-16
Boundary for River Rch & Prof#=Churchill River,Main            , 370
Up Type= 0
Dn Type= 1
Dn Known WS=-1.38778E-16
Boundary for River Rch & Prof#=Churchill River,Main            , 371
Up Type= 0
Dn Type= 1
Dn Known WS=-1.38778E-16
Boundary for River Rch & Prof#=Churchill River,Main            , 372
Up Type= 0
Dn Type= 1
Dn Known WS=-1.38778E-16
Boundary for River Rch & Prof#=Churchill River,Main            , 373
Up Type= 0
Dn Type= 1
Dn Known WS=-1.38778E-16
Boundary for River Rch & Prof#=Churchill River,Main            , 374
Up Type= 0
Dn Type= 1
Dn Known WS=-1.38778E-16
Boundary for River Rch & Prof#=Churchill River,Main            , 375
Up Type= 0
Dn Type= 1
Dn Known WS=-1.38778E-16
Boundary for River Rch & Prof#=Churchill River,Main            , 376
Up Type= 0
Dn Type= 1
Dn Known WS=-1.38778E-16
Boundary for River Rch & Prof#=Churchill River,Main            , 377
Up Type= 0
Dn Type= 1
Dn Known WS=-1.38778E-16
Boundary for River Rch & Prof#=Churchill River,Main            , 378
Up Type= 0
Dn Type= 1
Dn Known WS=-1.38778E-16
Boundary for River Rch & Prof#=Churchill River,Main            , 379
Up Type= 0
Dn Type= 1
Dn Known WS=-1.38778E-16
Boundary for River Rch & Prof#=Churchill River,Main            , 380
Up Type= 0
Dn Type= 1
Dn Known WS=-1.38778E-16
Boundary for River Rch & Prof#=Churchill River,Main            , 381
Up Type= 0
Dn Type= 1
Dn Known WS=-1.38778E-16
Boundary for River Rch & Prof#=Churchill River,Main            , 382
Up Type= 0
Dn Type= 1
Dn Known WS=-1.38778E-16
Boundary for River Rch & Prof#=Churchill River,Main            , 383
Up Type= 0
Dn Type= 1
Dn Known WS=-1.38778E-16
Boundary for River Rch & Prof#=Churchill River,Main            , 384
Up Type= 0
Dn Type= 1
Dn Known WS=-1.38778E-16
Boundary for River Rch & Prof#=Churchill River,Main            , 385
Up Type= 0
Dn Type= 1
Dn Known WS=-1.38778E-16
Boundary for River Rch & Prof#=Churchill River,Main            , 386
Up Type= 0
Dn Type= 1
Dn Known WS=0.1
Boundary for River Rch & Prof#=Churchill River,Main            , 387
Up Type= 0
Dn Type= 1
Dn Known WS=0.1
Boundary for River Rch & Prof#=Churchill River,Main            , 388
Up Type= 0
Dn Type= 1
Dn Known WS=0.1
Boundary for River Rch & Prof#=Churchill River,Main            , 389
Up Type= 0
Dn Type= 1
Dn Known WS=0.1
Boundary for River Rch & Prof#=Churchill River,Main            , 390
Up Type= 0
Dn Type= 1
Dn Known WS=0.1
Boundary for River Rch & Prof#=Churchill River,Main            , 391
Up Type= 0
Dn Type= 1
Dn Known WS=0.1
Boundary for River Rch & Prof#=Churchill River,Main            , 392
Up Type= 0
Dn Type= 1
Dn Known WS=0.1
Boundary for River Rch & Prof#=Churchill River,Main            , 393
Up Type= 0
Dn Type= 1
Dn Known WS=0.1
Boundary for River Rch & Prof#=Churchill River,Main            , 394
Up Type= 0
Dn Type= 1
Dn Known WS=0.1
Boundary for River Rch & Prof#=Churchill River,Main            , 395
Up Type= 0
Dn Type= 1
Dn Known WS=0.1
Boundary for River Rch & Prof#=Churchill River,Main            , 396
Up Type= 0
Dn Type= 1
Dn Known WS=0.1
Boundary for River Rch & Prof#=Churchill River,Main            , 397
Up Type= 0
Dn Type= 1
Dn Known WS=0.1
Boundary for River Rch & Prof#=Churchill River,Main            , 398
Up Type= 0
Dn Type= 1
Dn Known WS=0.1
Boundary for River Rch & Prof#=Churchill River,Main            , 399
Up Type= 0
Dn Type= 1
Dn Known WS=0.1
Boundary for River Rch & Prof#=Churchill River,Main            , 400
Up Type= 0
Dn Type= 1
Dn Known WS=0.1
Boundary for River Rch & Prof#=Churchill River,Main            , 401
Up Type= 0
Dn Type= 1
Dn Known WS=0.1
Boundary for River Rch & Prof#=Churchill River,Main            , 402
Up Type= 0
Dn Type= 1
Dn Known WS=0.1
Boundary for River Rch & Prof#=Churchill River,Main            , 403
Up Type= 0
Dn Type= 1
Dn Known WS=0.1
Boundary for River Rch & Prof#=Churchill River,Main            , 404
Up Type= 0
Dn Type= 1
Dn Known WS=0.1
Boundary for River Rch & Prof#=Churchill River,Main            , 405
Up Type= 0
Dn Type= 1
Dn Known WS=0.1
Boundary for River Rch & Prof#=Churchill River,Main            , 406
Up Type= 0
Dn Type= 1
Dn Known WS=0.1
Boundary for River Rch & Prof#=Churchill River,Main            , 407
Up Type= 0
Dn Type= 1
Dn Known WS=0.1
Boundary for River Rch & Prof#=Churchill River,Main            , 408
Up Type= 0
Dn Type= 1
Dn Known WS=0.1
Boundary for River Rch & Prof#=Churchill River,Main            , 409
Up Type= 0
Dn Type= 1
Dn Known WS=0.1
Boundary for River Rch & Prof#=Churchill River,Main            , 410
Up Type= 0
Dn Type= 1
Dn Known WS=0.1
Boundary for River Rch & Prof#=Churchill River,Main            , 411
Up Type= 0
Dn Type= 1
Dn Known WS=0.1
Boundary for River Rch & Prof#=Churchill River,Main            , 412
Up Type= 0
Dn Type= 1
Dn Known WS=0.1
Boundary for River Rch & Prof#=Churchill River,Main            , 413
Up Type= 0
Dn Type= 1
Dn Known WS=0.1
Boundary for River Rch & Prof#=Churchill River,Main            , 414
Up Type= 0
Dn Type= 1
Dn Known WS=0.1
Boundary for River Rch & Prof#=Churchill River,Main            , 415
Up Type= 0
Dn Type= 1
Dn Known WS=0.1
Boundary for River Rch & Prof#=Churchill River,Main            , 416
Up Type= 0
Dn Type= 1
Dn Known WS=0.1
Boundary for River Rch & Prof#=Churchill River,Main            , 417
Up Type= 0
Dn Type= 1
Dn Known WS=0.1
Boundary for River Rch & Prof#=Churchill River,Main            , 418
Up Type= 0
Dn Type= 1
Dn Known WS=0.1
Boundary for River Rch & Prof#=Churchill River,Main            , 419
Up Type= 0
Dn Type= 1
Dn Known WS=0.1
Boundary for River Rch & Prof#=Churchill River,Main            , 420
Up Type= 0
Dn Type= 1
Dn Known WS=0.1
Boundary for River Rch & Prof#=Churchill River,Main            , 421
Up Type= 0
Dn Type= 1
Dn Known WS=0.2
Boundary for River Rch & Prof#=Churchill River,Main            , 422
Up Type= 0
Dn Type= 1
Dn Known WS=0.2
Boundary for River Rch & Prof#=Churchill River,Main            , 423
Up Type= 0
Dn Type= 1
Dn Known WS=0.2
Boundary for River Rch & Prof#=Churchill River,Main            , 424
Up Type= 0
Dn Type= 1
Dn Known WS=0.2
Boundary for River Rch & Prof#=Churchill River,Main            , 425
Up Type= 0
Dn Type= 1
Dn Known WS=0.2
Boundary for River Rch & Prof#=Churchill River,Main            , 426
Up Type= 0
Dn Type= 1
Dn Known WS=0.2
Boundary for River Rch & Prof#=Churchill River,Main            , 427
Up Type= 0
Dn Type= 1
Dn Known WS=0.2
Boundary for River Rch & Prof#=Churchill River,Main            , 428
Up Type= 0
Dn Type= 1
Dn Known WS=0.2
Boundary for River Rch & Prof#=Churchill River,Main            , 429
Up Type= 0
Dn Type= 1
Dn Known WS=0.2
Boundary for River Rch & Prof#=Churchill River,Main            , 430
Up Type= 0
Dn Type= 1
Dn Known WS=0.2
Boundary for River Rch & Prof#=Churchill River,Main            , 431
Up Type= 0
Dn Type= 1
Dn Known WS=0.2
Boundary for River Rch & Prof#=Churchill River,Main            , 432
Up Type= 0
Dn Type= 1
Dn Known WS=0.2
Boundary for River Rch & Prof#=Churchill River,Main            , 433
Up Type= 0
Dn Type= 1
Dn Known WS=0.2
Boundary for River Rch & Prof#=Churchill River,Main            , 434
Up Type= 0
Dn Type= 1
Dn Known WS=0.2
Boundary for River Rch & Prof#=Churchill River,Main            , 435
Up Type= 0
Dn Type= 1
Dn Known WS=0.2
Boundary for River Rch & Prof#=Churchill River,Main            , 436
Up Type= 0
Dn Type= 1
Dn Known WS=0.2
Boundary for River Rch & Prof#=Churchill River,Main            , 437
Up Type= 0
Dn Type= 1
Dn Known WS=0.2
Boundary for River Rch & Prof#=Churchill River,Main            , 438
Up Type= 0
Dn Type= 1
Dn Known WS=0.2
Boundary for River Rch & Prof#=Churchill River,Main            , 439
Up Type= 0
Dn Type= 1
Dn Known WS=0.2
Boundary for River Rch & Prof#=Churchill River,Main            , 440
Up Type= 0
Dn Type= 1
Dn Known WS=0.2
Boundary for River Rch & Prof#=Churchill River,Main            , 441
Up Type= 0
Dn Type= 1
Dn Known WS=0.2
Boundary for River Rch & Prof#=Churchill River,Main            , 442
Up Type= 0
Dn Type= 1
Dn Known WS=0.2
Boundary for River Rch & Prof#=Churchill River,Main            , 443
Up Type= 0
Dn Type= 1
Dn Known WS=0.2
Boundary for River Rch & Prof#=Churchill River,Main            , 444
Up Type= 0
Dn Type= 1
Dn Known WS=0.2
Boundary for River Rch & Prof#=Churchill River,Main            , 445
Up Type= 0
Dn Type= 1
Dn Known WS=0.2
Boundary for River Rch & Prof#=Churchill River,Main            , 446
Up Type= 0
Dn Type= 1
Dn Known WS=0.2
Boundary for River Rch & Prof#=Churchill River,Main            , 447
Up Type= 0
Dn Type= 1
Dn Known WS=0.2
Boundary for River Rch & Prof#=Churchill River,Main            , 448
Up Type= 0
Dn Type= 1
Dn Known WS=0.2
Boundary for River Rch & Prof#=Churchill River,Main            , 449
Up Type= 0
Dn Type= 1
Dn Known WS=0.2
Boundary for River Rch & Prof#=Churchill River,Main            , 450
Up Type= 0
Dn Type= 1
Dn Known WS=0.2
Boundary for River Rch & Prof#=Churchill River,Main            , 451
Up Type= 0
Dn Type= 1
Dn Known WS=0.2
Boundary for River Rch & Prof#=Churchill River,Main            , 452
Up Type= 0
Dn Type= 1
Dn Known WS=0.2
Boundary for River Rch & Prof#=Churchill River,Main            , 453
Up Type= 0
Dn Type= 1
Dn Known WS=0.2
Boundary for River Rch & Prof#=Churchill River,Main            , 454
Up Type= 0
Dn Type= 1
Dn Known WS=0.2
Boundary for River Rch & Prof#=Churchill River,Main            , 455
Up Type= 0
Dn Type= 1
Dn Known WS=0.2
Boundary for River Rch & Prof#=Churchill River,Main            , 456
Up Type= 0
Dn Type= 1
Dn Known WS=0.3
Boundary for River Rch & Prof#=Churchill River,Main            , 457
Up Type= 0
Dn Type= 1
Dn Known WS=0.3
Boundary for River Rch & Prof#=Churchill River,Main            , 458
Up Type= 0
Dn Type= 1
Dn Known WS=0.3
Boundary for River Rch & Prof#=Churchill River,Main            , 459
Up Type= 0
Dn Type= 1
Dn Known WS=0.3
Boundary for River Rch & Prof#=Churchill River,Main            , 460
Up Type= 0
Dn Type= 1
Dn Known WS=0.3
Boundary for River Rch & Prof#=Churchill River,Main            , 461
Up Type= 0
Dn Type= 1
Dn Known WS=0.3
Boundary for River Rch & Prof#=Churchill River,Main            , 462
Up Type= 0
Dn Type= 1
Dn Known WS=0.3
Boundary for River Rch & Prof#=Churchill River,Main            , 463
Up Type= 0
Dn Type= 1
Dn Known WS=0.3
Boundary for River Rch & Prof#=Churchill River,Main            , 464
Up Type= 0
Dn Type= 1
Dn Known WS=0.3
Boundary for River Rch & Prof#=Churchill River,Main            , 465
Up Type= 0
Dn Type= 1
Dn Known WS=0.3
Boundary for River Rch & Prof#=Churchill River,Main            , 466
Up Type= 0
Dn Type= 1
Dn Known WS=0.3
Boundary for River Rch & Prof#=Churchill River,Main            , 467
Up Type= 0
Dn Type= 1
Dn Known WS=0.3
Boundary for River Rch & Prof#=Churchill River,Main            , 468
Up Type= 0
Dn Type= 1
Dn Known WS=0.3
Boundary for River Rch & Prof#=Churchill River,Main            , 469
Up Type= 0
Dn Type= 1
Dn Known WS=0.3
Boundary for River Rch & Prof#=Churchill River,Main            , 470
Up Type= 0
Dn Type= 1
Dn Known WS=0.3
Boundary for River Rch & Prof#=Churchill River,Main            , 471
Up Type= 0
Dn Type= 1
Dn Known WS=0.3
Boundary for River Rch & Prof#=Churchill River,Main            , 472
Up Type= 0
Dn Type= 1
Dn Known WS=0.3
Boundary for River Rch & Prof#=Churchill River,Main            , 473
Up Type= 0
Dn Type= 1
Dn Known WS=0.3
Boundary for River Rch & Prof#=Churchill River,Main            , 474
Up Type= 0
Dn Type= 1
Dn Known WS=0.3
Boundary for River Rch & Prof#=Churchill River,Main            , 475
Up Type= 0
Dn Type= 1
Dn Known WS=0.3
Boundary for River Rch & Prof#=Churchill River,Main            , 476
Up Type= 0
Dn Type= 1
Dn Known WS=0.3
Boundary for River Rch & Prof#=Churchill River,Main            , 477
Up Type= 0
Dn Type= 1
Dn Known WS=0.3
Boundary for River Rch & Prof#=Churchill River,Main            , 478
Up Type= 0
Dn Type= 1
Dn Known WS=0.3
Boundary for River Rch & Prof#=Churchill River,Main            , 479
Up Type= 0
Dn Type= 1
Dn Known WS=0.3
Boundary for River Rch & Prof#=Churchill River,Main            , 480
Up Type= 0
Dn Type= 1
Dn Known WS=0.3
Boundary for River Rch & Prof#=Churchill River,Main            , 481
Up Type= 0
Dn Type= 1
Dn Known WS=0.3
Boundary for River Rch & Prof#=Churchill River,Main            , 482
Up Type= 0
Dn Type= 1
Dn Known WS=0.3
Boundary for River Rch & Prof#=Churchill River,Main            , 483
Up Type= 0
Dn Type= 1
Dn Known WS=0.3
Boundary for River Rch & Prof#=Churchill River,Main            , 484
Up Type= 0
Dn Type= 1
Dn Known WS=0.3
Boundary for River Rch & Prof#=Churchill River,Main            , 485
Up Type= 0
Dn Type= 1
Dn Known WS=0.3
Boundary for River Rch & Prof#=Churchill River,Main            , 486
Up Type= 0
Dn Type= 1
Dn Known WS=0.3
Boundary for River Rch & Prof#=Churchill River,Main            , 487
Up Type= 0
Dn Type= 1
Dn Known WS=0.3
Boundary for River Rch & Prof#=Churchill River,Main            , 488
Up Type= 0
Dn Type= 1
Dn Known WS=0.3
Boundary for River Rch & Prof#=Churchill River,Main            , 489
Up Type= 0
Dn Type= 1
Dn Known WS=0.3
Boundary for River Rch & Prof#=Churchill River,Main            , 490
Up Type= 0
Dn Type= 1
Dn Known WS=0.3
Boundary for River Rch & Prof#=Churchill River,Main            , 491
Up Type= 0
Dn Type= 1
Dn Known WS=0.4
Boundary for River Rch & Prof#=Churchill River,Main            , 492
Up Type= 0
Dn Type= 1
Dn Known WS=0.4
Boundary for River Rch & Prof#=Churchill River,Main            , 493
Up Type= 0
Dn Type= 1
Dn Known WS=0.4
Boundary for River Rch & Prof#=Churchill River,Main            , 494
Up Type= 0
Dn Type= 1
Dn Known WS=0.4
Boundary for River Rch & Prof#=Churchill River,Main            , 495
Up Type= 0
Dn Type= 1
Dn Known WS=0.4
Boundary for River Rch & Prof#=Churchill River,Main            , 496
Up Type= 0
Dn Type= 1
Dn Known WS=0.4
Boundary for River Rch & Prof#=Churchill River,Main            , 497
Up Type= 0
Dn Type= 1
Dn Known WS=0.4
Boundary for River Rch & Prof#=Churchill River,Main            , 498
Up Type= 0
Dn Type= 1
Dn Known WS=0.4
Boundary for River Rch & Prof#=Churchill River,Main            , 499
Up Type= 0
Dn Type= 1
Dn Known WS=0.4
Boundary for River Rch & Prof#=Churchill River,Main            , 500
Up Type= 0
Dn Type= 1
Dn Known WS=0.4
Boundary for River Rch & Prof#=Churchill River,Main            , 501
Up Type= 0
Dn Type= 1
Dn Known WS=0.4
Boundary for River Rch & Prof#=Churchill River,Main            , 502
Up Type= 0
Dn Type= 1
Dn Known WS=0.4
Boundary for River Rch & Prof#=Churchill River,Main            , 503
Up Type= 0
Dn Type= 1
Dn Known WS=0.4
Boundary for River Rch & Prof#=Churchill River,Main            , 504
Up Type= 0
Dn Type= 1
Dn Known WS=0.4
Boundary for River Rch & Prof#=Churchill River,Main            , 505
Up Type= 0
Dn Type= 1
Dn Known WS=0.4
Boundary for River Rch & Prof#=Churchill River,Main            , 506
Up Type= 0
Dn Type= 1
Dn Known WS=0.4
Boundary for River Rch & Prof#=Churchill River,Main            , 507
Up Type= 0
Dn Type= 1
Dn Known WS=0.4
Boundary for River Rch & Prof#=Churchill River,Main            , 508
Up Type= 0
Dn Type= 1
Dn Known WS=0.4
Boundary for River Rch & Prof#=Churchill River,Main            , 509
Up Type= 0
Dn Type= 1
Dn Known WS=0.4
Boundary for River Rch & Prof#=Churchill River,Main            , 510
Up Type= 0
Dn Type= 1
Dn Known WS=0.4
Boundary for River Rch & Prof#=Churchill River,Main            , 511
Up Type= 0
Dn Type= 1
Dn Known WS=0.4
Boundary for River Rch & Prof#=Churchill River,Main            , 512
Up Type= 0
Dn Type= 1
Dn Known WS=0.4
Boundary for River Rch & Prof#=Churchill River,Main            , 513
Up Type= 0
Dn Type= 1
Dn Known WS=0.4
Boundary for River Rch & Prof#=Churchill River,Main            , 514
Up Type= 0
Dn Type= 1
Dn Known WS=0.4
Boundary for River Rch & Prof#=Churchill River,Main            , 515
Up Type= 0
Dn Type= 1
Dn Known WS=0.4
Boundary for River Rch & Prof#=Churchill River,Main            , 516
Up Type= 0
Dn Type= 1
Dn Known WS=0.4
Boundary for River Rch & Prof#=Churchill River,Main            , 517
Up Type= 0
Dn Type= 1
Dn Known WS=0.4
Boundary for River Rch & Prof#=Churchill River,Main            , 518
Up Type= 0
Dn Type= 1
Dn Known WS=0.4
Boundary for River Rch & Prof#=Churchill River,Main            , 519
Up Type= 0
Dn Type= 1
Dn Known WS=0.4
Boundary for River Rch & Prof#=Churchill River,Main            , 520
Up Type= 0
Dn Type= 1
Dn Known WS=0.4
Boundary for River Rch & Prof#=Churchill River,Main            , 521
Up Type= 0
Dn Type= 1
Dn Known WS=0.4
Boundary for River Rch & Prof#=Churchill River,Main            , 522
Up Type= 0
Dn Type= 1
Dn Known WS=0.4
Boundary for River Rch & Prof#=Churchill River,Main            , 523
Up Type= 0
Dn Type= 1
Dn Known WS=0.4
Boundary for River Rch & Prof#=Churchill River,Main            , 524
Up Type= 0
Dn Type= 1
Dn Known WS=0.4
Boundary for River Rch & Prof#=Churchill River,Main            , 525
Up Type= 0
Dn Type= 1
Dn Known WS=0.4
Boundary for River Rch & Prof#=Churchill River,Main            , 526
Up Type= 0
Dn Type= 1
Dn Known WS=0.5
Boundary for River Rch & Prof#=Churchill River,Main            , 527
Up Type= 0
Dn Type= 1
Dn Known WS=0.5
Boundary for River Rch & Prof#=Churchill River,Main            , 528
Up Type= 0
Dn Type= 1
Dn Known WS=0.5
Boundary for River Rch & Prof#=Churchill River,Main            , 529
Up Type= 0
Dn Type= 1
Dn Known WS=0.5
Boundary for River Rch & Prof#=Churchill River,Main            , 530
Up Type= 0
Dn Type= 1
Dn Known WS=0.5
Boundary for River Rch & Prof#=Churchill River,Main            , 531
Up Type= 0
Dn Type= 1
Dn Known WS=0.5
Boundary for River Rch & Prof#=Churchill River,Main            , 532
Up Type= 0
Dn Type= 1
Dn Known WS=0.5
Boundary for River Rch & Prof#=Churchill River,Main            , 533
Up Type= 0
Dn Type= 1
Dn Known WS=0.5
Boundary for River Rch & Prof#=Churchill River,Main            , 534
Up Type= 0
Dn Type= 1
Dn Known WS=0.5
Boundary for River Rch & Prof#=Churchill River,Main            , 535
Up Type= 0
Dn Type= 1
Dn Known WS=0.5
Boundary for River Rch & Prof#=Churchill River,Main            , 536
Up Type= 0
Dn Type= 1
Dn Known WS=0.5
Boundary for River Rch & Prof#=Churchill River,Main            , 537
Up Type= 0
Dn Type= 1
Dn Known WS=0.5
Boundary for River Rch & Prof#=Churchill River,Main            , 538
Up Type= 0
Dn Type= 1
Dn Known WS=0.5
Boundary for River Rch & Prof#=Churchill River,Main            , 539
Up Type= 0
Dn Type= 1
Dn Known WS=0.5
Boundary for River Rch & Prof#=Churchill River,Main            , 540
Up Type= 0
Dn Type= 1
Dn Known WS=0.5
Boundary for River Rch & Prof#=Churchill River,Main            , 541
Up Type= 0
Dn Type= 1
Dn Known WS=0.5
Boundary for River Rch & Prof#=Churchill River,Main            , 542
Up Type= 0
Dn Type= 1
Dn Known WS=0.5
Boundary for River Rch & Prof#=Churchill River,Main            , 543
Up Type= 0
Dn Type= 1
Dn Known WS=0.5
Boundary for River Rch & Prof#=Churchill River,Main            , 544
Up Type= 0
Dn Type= 1
Dn Known WS=0.5
Boundary for River Rch & Prof#=Churchill River,Main            , 545
Up Type= 0
Dn Type= 1
Dn Known WS=0.5
Boundary for River Rch & Prof#=Churchill River,Main            , 546
Up Type= 0
Dn Type= 1
Dn Known WS=0.5
Boundary for River Rch & Prof#=Churchill River,Main            , 547
Up Type= 0
Dn Type= 1
Dn Known WS=0.5
Boundary for River Rch & Prof#=Churchill River,Main            , 548
Up Type= 0
Dn Type= 1
Dn Known WS=0.5
Boundary for River Rch & Prof#=Churchill River,Main            , 549
Up Type= 0
Dn Type= 1
Dn Known WS=0.5
Boundary for River Rch & Prof#=Churchill River,Main            , 550
Up Type= 0
Dn Type= 1
Dn Known WS=0.5
Boundary for River Rch & Prof#=Churchill River,Main            , 551
Up Type= 0
Dn Type= 1
Dn Known WS=0.5
Boundary for River Rch & Prof#=Churchill River,Main            , 552
Up Type= 0
Dn Type= 1
Dn Known WS=0.5
Boundary for River Rch & Prof#=Churchill River,Main            , 553
Up Type= 0
Dn Type= 1
Dn Known WS=0.5
Boundary for River Rch & Prof#=Churchill River,Main            , 554
Up Type= 0
Dn Type= 1
Dn Known WS=0.5
Boundary for River Rch & Prof#=Churchill River,Main            , 555
Up Type= 0
Dn Type= 1
Dn Known WS=0.5
Boundary for River Rch & Prof#=Churchill River,Main            , 556
Up Type= 0
Dn Type= 1
Dn Known WS=0.5
Boundary for River Rch & Prof#=Churchill River,Main            , 557
Up Type= 0
Dn Type= 1
Dn Known WS=0.5
Boundary for River Rch & Prof#=Churchill River,Main            , 558
Up Type= 0
Dn Type= 1
Dn Known WS=0.5
Boundary for River Rch & Prof#=Churchill River,Main            , 559
Up Type= 0
Dn Type= 1
Dn Known WS=0.5
Boundary for River Rch & Prof#=Churchill River,Main            , 560
Up Type= 0
Dn Type= 1
Dn Known WS=0.5
Boundary for River Rch & Prof#=Churchill River,Main            , 561
Up Type= 0
Dn Type= 1
Dn Known WS=0.6
Boundary for River Rch & Prof#=Churchill River,Main            , 562
Up Type= 0
Dn Type= 1
Dn Known WS=0.6
Boundary for River Rch & Prof#=Churchill River,Main            , 563
Up Type= 0
Dn Type= 1
Dn Known WS=0.6
Boundary for River Rch & Prof#=Churchill River,Main            , 564
Up Type= 0
Dn Type= 1
Dn Known WS=0.6
Boundary for River Rch & Prof#=Churchill River,Main            , 565
Up Type= 0
Dn Type= 1
Dn Known WS=0.6
Boundary for River Rch & Prof#=Churchill River,Main            , 566
Up Type= 0
Dn Type= 1
Dn Known WS=0.6
Boundary for River Rch & Prof#=Churchill River,Main            , 567
Up Type= 0
Dn Type= 1
Dn Known WS=0.6
Boundary for River Rch & Prof#=Churchill River,Main            , 568
Up Type= 0
Dn Type= 1
Dn Known WS=0.6
Boundary for River Rch & Prof#=Churchill River,Main            , 569
Up Type= 0
Dn Type= 1
Dn Known WS=0.6
Boundary for River Rch & Prof#=Churchill River,Main            , 570
Up Type= 0
Dn Type= 1
Dn Known WS=0.6
Boundary for River Rch & Prof#=Churchill River,Main            , 571
Up Type= 0
Dn Type= 1
Dn Known WS=0.6
Boundary for River Rch & Prof#=Churchill River,Main            , 572
Up Type= 0
Dn Type= 1
Dn Known WS=0.6
Boundary for River Rch & Prof#=Churchill River,Main            , 573
Up Type= 0
Dn Type= 1
Dn Known WS=0.6
Boundary for River Rch & Prof#=Churchill River,Main            , 574
Up Type= 0
Dn Type= 1
Dn Known WS=0.6
Boundary for River Rch & Prof#=Churchill River,Main            , 575
Up Type= 0
Dn Type= 1
Dn Known WS=0.6
Boundary for River Rch & Prof#=Churchill River,Main            , 576
Up Type= 0
Dn Type= 1
Dn Known WS=0.6
Boundary for River Rch & Prof#=Churchill River,Main            , 577
Up Type= 0
Dn Type= 1
Dn Known WS=0.6
Boundary for River Rch & Prof#=Churchill River,Main            , 578
Up Type= 0
Dn Type= 1
Dn Known WS=0.6
Boundary for River Rch & Prof#=Churchill River,Main            , 579
Up Type= 0
Dn Type= 1
Dn Known WS=0.6
Boundary for River Rch & Prof#=Churchill River,Main            , 580
Up Type= 0
Dn Type= 1
Dn Known WS=0.6
Boundary for River Rch & Prof#=Churchill River,Main            , 581
Up Type= 0
Dn Type= 1
Dn Known WS=0.6
Boundary for River Rch & Prof#=Churchill River,Main            , 582
Up Type= 0
Dn Type= 1
Dn Known WS=0.6
Boundary for River Rch & Prof#=Churchill River,Main            , 583
Up Type= 0
Dn Type= 1
Dn Known WS=0.6
Boundary for River Rch & Prof#=Churchill River,Main            , 584
Up Type= 0
Dn Type= 1
Dn Known WS=0.6
Boundary for River Rch & Prof#=Churchill River,Main            , 585
Up Type= 0
Dn Type= 1
Dn Known WS=0.6
Boundary for River Rch & Prof#=Churchill River,Main            , 586
Up Type= 0
Dn Type= 1
Dn Known WS=0.6
Boundary for River Rch & Prof#=Churchill River,Main            , 587
Up Type= 0
Dn Type= 1
Dn Known WS=0.6
Boundary for River Rch & Prof#=Churchill River,Main            , 588
Up Type= 0
Dn Type= 1
Dn Known WS=0.6
Boundary for River Rch & Prof#=Churchill River,Main            , 589
Up Type= 0
Dn Type= 1
Dn Known WS=0.6
Boundary for River Rch & Prof#=Churchill River,Main            , 590
Up Type= 0
Dn Type= 1
Dn Known WS=0.6
Boundary for River Rch & Prof#=Churchill River,Main            , 591
Up Type= 0
Dn Type= 1
Dn Known WS=0.6
Boundary for River Rch & Prof#=Churchill River,Main            , 592
Up Type= 0
Dn Type= 1
Dn Known WS=0.6
Boundary for River Rch & Prof#=Churchill River,Main            , 593
Up Type= 0
Dn Type= 1
Dn Known WS=0.6
Boundary for River Rch & Prof#=Churchill River,Main            , 594
Up Type= 0
Dn Type= 1
Dn Known WS=0.6
Boundary for River Rch & Prof#=Churchill River,Main            , 595
Up Type= 0
Dn Type= 1
Dn Known WS=0.6
Boundary for River Rch & Prof#=Churchill River,Main            , 596
Up Type= 0
Dn Type= 1
Dn Known WS=0.7
Boundary for River Rch & Prof#=Churchill River,Main            , 597
Up Type= 0
Dn Type= 1
Dn Known WS=0.7
Boundary for River Rch & Prof#=Churchill River,Main            , 598
Up Type= 0
Dn Type= 1
Dn Known WS=0.7
Boundary for River Rch & Prof#=Churchill River,Main            , 599
Up Type= 0
Dn Type= 1
Dn Known WS=0.7
Boundary for River Rch & Prof#=Churchill River,Main            , 600
Up Type= 0
Dn Type= 1
Dn Known WS=0.7
Boundary for River Rch & Prof#=Churchill River,Main            , 601
Up Type= 0
Dn Type= 1
Dn Known WS=0.7
Boundary for River Rch & Prof#=Churchill River,Main            , 602
Up Type= 0
Dn Type= 1
Dn Known WS=0.7
Boundary for River Rch & Prof#=Churchill River,Main            , 603
Up Type= 0
Dn Type= 1
Dn Known WS=0.7
Boundary for River Rch & Prof#=Churchill River,Main            , 604
Up Type= 0
Dn Type= 1
Dn Known WS=0.7
Boundary for River Rch & Prof#=Churchill River,Main            , 605
Up Type= 0
Dn Type= 1
Dn Known WS=0.7
Boundary for River Rch & Prof#=Churchill River,Main            , 606
Up Type= 0
Dn Type= 1
Dn Known WS=0.7
Boundary for River Rch & Prof#=Churchill River,Main            , 607
Up Type= 0
Dn Type= 1
Dn Known WS=0.7
Boundary for River Rch & Prof#=Churchill River,Main            , 608
Up Type= 0
Dn Type= 1
Dn Known WS=0.7
Boundary for River Rch & Prof#=Churchill River,Main            , 609
Up Type= 0
Dn Type= 1
Dn Known WS=0.7
Boundary for River Rch & Prof#=Churchill River,Main            , 610
Up Type= 0
Dn Type= 1
Dn Known WS=0.7
Boundary for River Rch & Prof#=Churchill River,Main            , 611
Up Type= 0
Dn Type= 1
Dn Known WS=0.7
Boundary for River Rch & Prof#=Churchill River,Main            , 612
Up Type= 0
Dn Type= 1
Dn Known WS=0.7
Boundary for River Rch & Prof#=Churchill River,Main            , 613
Up Type= 0
Dn Type= 1
Dn Known WS=0.7
Boundary for River Rch & Prof#=Churchill River,Main            , 614
Up Type= 0
Dn Type= 1
Dn Known WS=0.7
Boundary for River Rch & Prof#=Churchill River,Main            , 615
Up Type= 0
Dn Type= 1
Dn Known WS=0.7
Boundary for River Rch & Prof#=Churchill River,Main            , 616
Up Type= 0
Dn Type= 1
Dn Known WS=0.7
Boundary for River Rch & Prof#=Churchill River,Main            , 617
Up Type= 0
Dn Type= 1
Dn Known WS=0.7
Boundary for River Rch & Prof#=Churchill River,Main            , 618
Up Type= 0
Dn Type= 1
Dn Known WS=0.7
Boundary for River Rch & Prof#=Churchill River,Main            , 619
Up Type= 0
Dn Type= 1
Dn Known WS=0.7
Boundary for River Rch & Prof#=Churchill River,Main            , 620
Up Type= 0
Dn Type= 1
Dn Known WS=0.7
Boundary for River Rch & Prof#=Churchill River,Main            , 621
Up Type= 0
Dn Type= 1
Dn Known WS=0.7
Boundary for River Rch & Prof#=Churchill River,Main            , 622
Up Type= 0
Dn Type= 1
Dn Known WS=0.7
Boundary for River Rch & Prof#=Churchill River,Main            , 623
Up Type= 0
Dn Type= 1
Dn Known WS=0.7
Boundary for River Rch & Prof#=Churchill River,Main            , 624
Up Type= 0
Dn Type= 1
Dn Known WS=0.7
Boundary for River Rch & Prof#=Churchill River,Main            , 625
Up Type= 0
Dn Type= 1
Dn Known WS=0.7
Boundary for River Rch & Prof#=Churchill River,Main            , 626
Up Type= 0
Dn Type= 1
Dn Known WS=0.7
Boundary for River Rch & Prof#=Churchill River,Main            , 627
Up Type= 0
Dn Type= 1
Dn Known WS=0.7
Boundary for River Rch & Prof#=Churchill River,Main            , 628
Up Type= 0
Dn Type= 1
Dn Known WS=0.7
Boundary for River Rch & Prof#=Churchill River,Main            , 629
Up Type= 0
Dn Type= 1
Dn Known WS=0.7
Boundary for River Rch & Prof#=Churchill River,Main            , 630
Up Type= 0
Dn Type= 1
Dn Known WS=0.7
Boundary for River Rch & Prof#=Churchill River,Main            , 631
Up Type= 0
Dn Type= 1
Dn Known WS=0.8
Boundary for River Rch & Prof#=Churchill River,Main            , 632
Up Type= 0
Dn Type= 1
Dn Known WS=0.8
Boundary for River Rch & Prof#=Churchill River,Main            , 633
Up Type= 0
Dn Type= 1
Dn Known WS=0.8
Boundary for River Rch & Prof#=Churchill River,Main            , 634
Up Type= 0
Dn Type= 1
Dn Known WS=0.8
Boundary for River Rch & Prof#=Churchill River,Main            , 635
Up Type= 0
Dn Type= 1
Dn Known WS=0.8
Boundary for River Rch & Prof#=Churchill River,Main            , 636
Up Type= 0
Dn Type= 1
Dn Known WS=0.8
Boundary for River Rch & Prof#=Churchill River,Main            , 637
Up Type= 0
Dn Type= 1
Dn Known WS=0.8
Boundary for River Rch & Prof#=Churchill River,Main            , 638
Up Type= 0
Dn Type= 1
Dn Known WS=0.8
Boundary for River Rch & Prof#=Churchill River,Main            , 639
Up Type= 0
Dn Type= 1
Dn Known WS=0.8
Boundary for River Rch & Prof#=Churchill River,Main            , 640
Up Type= 0
Dn Type= 1
Dn Known WS=0.8
Boundary for River Rch & Prof#=Churchill River,Main            , 641
Up Type= 0
Dn Type= 1
Dn Known WS=0.8
Boundary for River Rch & Prof#=Churchill River,Main            , 642
Up Type= 0
Dn Type= 1
Dn Known WS=0.8
Boundary for River Rch & Prof#=Churchill River,Main            , 643
Up Type= 0
Dn Type= 1
Dn Known WS=0.8
Boundary for River Rch & Prof#=Churchill River,Main            , 644
Up Type= 0
Dn Type= 1
Dn Known WS=0.8
Boundary for River Rch & Prof#=Churchill River,Main            , 645
Up Type= 0
Dn Type= 1
Dn Known WS=0.8
Boundary for River Rch & Prof#=Churchill River,Main            , 646
Up Type= 0
Dn Type= 1
Dn Known WS=0.8
Boundary for River Rch & Prof#=Churchill River,Main            , 647
Up Type= 0
Dn Type= 1
Dn Known WS=0.8
Boundary for River Rch & Prof#=Churchill River,Main            , 648
Up Type= 0
Dn Type= 1
Dn Known WS=0.8
Boundary for River Rch & Prof#=Churchill River,Main            , 649
Up Type= 0
Dn Type= 1
Dn Known WS=0.8
Boundary for River Rch & Prof#=Churchill River,Main            , 650
Up Type= 0
Dn Type= 1
Dn Known WS=0.8
Boundary for River Rch & Prof#=Churchill River,Main            , 651
Up Type= 0
Dn Type= 1
Dn Known WS=0.8
Boundary for River Rch & Prof#=Churchill River,Main            , 652
Up Type= 0
Dn Type= 1
Dn Known WS=0.8
Boundary for River Rch & Prof#=Churchill River,Main            , 653
Up Type= 0
Dn Type= 1
Dn Known WS=0.8
Boundary for River Rch & Prof#=Churchill River,Main            , 654
Up Type= 0
Dn Type= 1
Dn Known WS=0.8
Boundary for River Rch & Prof#=Churchill River,Main            , 655
Up Type= 0
Dn Type= 1
Dn Known WS=0.8
Boundary for River Rch & Prof#=Churchill River,Main            , 656
Up Type= 0
Dn Type= 1
Dn Known WS=0.8
Boundary for River Rch & Prof#=Churchill River,Main            , 657
Up Type= 0
Dn Type= 1
Dn Known WS=0.8
Boundary for River Rch & Prof#=Churchill River,Main            , 658
Up Type= 0
Dn Type= 1
Dn Known WS=0.8
Boundary for River Rch & Prof#=Churchill River,Main            , 659
Up Type= 0
Dn Type= 1
Dn Known WS=0.8
Boundary for River Rch & Prof#=Churchill River,Main            , 660
Up Type= 0
Dn Type= 1
Dn Known WS=0.8
Boundary for River Rch & Prof#=Churchill River,Main            , 661
Up Type= 0
Dn Type= 1
Dn Known WS=0.8
Boundary for River Rch & Prof#=Churchill River,Main            , 662
Up Type= 0
Dn Type= 1
Dn Known WS=0.8
Boundary for River Rch & Prof#=Churchill River,Main            , 663
Up Type= 0
Dn Type= 1
Dn Known WS=0.8
Boundary for River Rch & Prof#=Churchill River,Main            , 664
Up Type= 0
Dn Type= 1
Dn Known WS=0.8
Boundary for River Rch & Prof#=Churchill River,Main            , 665
Up Type= 0
Dn Type= 1
Dn Known WS=0.8
Boundary for River Rch & Prof#=Churchill River,Main            , 666
Up Type= 0
Dn Type= 1
Dn Known WS=0.9
Boundary for River Rch & Prof#=Churchill River,Main            , 667
Up Type= 0
Dn Type= 1
Dn Known WS=0.9
Boundary for River Rch & Prof#=Churchill River,Main            , 668
Up Type= 0
Dn Type= 1
Dn Known WS=0.9
Boundary for River Rch & Prof#=Churchill River,Main            , 669
Up Type= 0
Dn Type= 1
Dn Known WS=0.9
Boundary for River Rch & Prof#=Churchill River,Main            , 670
Up Type= 0
Dn Type= 1
Dn Known WS=0.9
Boundary for River Rch & Prof#=Churchill River,Main            , 671
Up Type= 0
Dn Type= 1
Dn Known WS=0.9
Boundary for River Rch & Prof#=Churchill River,Main            , 672
Up Type= 0
Dn Type= 1
Dn Known WS=0.9
Boundary for River Rch & Prof#=Churchill River,Main            , 673
Up Type= 0
Dn Type= 1
Dn Known WS=0.9
Boundary for River Rch & Prof#=Churchill River,Main            , 674
Up Type= 0
Dn Type= 1
Dn Known WS=0.9
Boundary for River Rch & Prof#=Churchill River,Main            , 675
Up Type= 0
Dn Type= 1
Dn Known WS=0.9
Boundary for River Rch & Prof#=Churchill River,Main            , 676
Up Type= 0
Dn Type= 1
Dn Known WS=0.9
Boundary for River Rch & Prof#=Churchill River,Main            , 677
Up Type= 0
Dn Type= 1
Dn Known WS=0.9
Boundary for River Rch & Prof#=Churchill River,Main            , 678
Up Type= 0
Dn Type= 1
Dn Known WS=0.9
Boundary for River Rch & Prof#=Churchill River,Main            , 679
Up Type= 0
Dn Type= 1
Dn Known WS=0.9
Boundary for River Rch & Prof#=Churchill River,Main            , 680
Up Type= 0
Dn Type= 1
Dn Known WS=0.9
Boundary for River Rch & Prof#=Churchill River,Main            , 681
Up Type= 0
Dn Type= 1
Dn Known WS=0.9
Boundary for River Rch & Prof#=Churchill River,Main            , 682
Up Type= 0
Dn Type= 1
Dn Known WS=0.9
Boundary for River Rch & Prof#=Churchill River,Main            , 683
Up Type= 0
Dn Type= 1
Dn Known WS=0.9
Boundary for River Rch & Prof#=Churchill River,Main            , 684
Up Type= 0
Dn Type= 1
Dn Known WS=0.9
Boundary for River Rch & Prof#=Churchill River,Main            , 685
Up Type= 0
Dn Type= 1
Dn Known WS=0.9
Boundary for River Rch & Prof#=Churchill River,Main            , 686
Up Type= 0
Dn Type= 1
Dn Known WS=0.9
Boundary for River Rch & Prof#=Churchill River,Main            , 687
Up Type= 0
Dn Type= 1
Dn Known WS=0.9
Boundary for River Rch & Prof#=Churchill River,Main            , 688
Up Type= 0
Dn Type= 1
Dn Known WS=0.9
Boundary for River Rch & Prof#=Churchill River,Main            , 689
Up Type= 0
Dn Type= 1
Dn Known WS=0.9
Boundary for River Rch & Prof#=Churchill River,Main            , 690
Up Type= 0
Dn Type= 1
Dn Known WS=0.9
Boundary for River Rch & Prof#=Churchill River,Main            , 691
Up Type= 0
Dn Type= 1
Dn Known WS=0.9
Boundary for River Rch & Prof#=Churchill River,Main            , 692
Up Type= 0
Dn Type= 1
Dn Known WS=0.9
Boundary for River Rch & Prof#=Churchill River,Main            , 693
Up Type= 0
Dn Type= 1
Dn Known WS=0.9
Boundary for River Rch & Prof#=Churchill River,Main            , 694
Up Type= 0
Dn Type= 1
Dn Known WS=0.9
Boundary for River Rch & Prof#=Churchill River,Main            , 695
Up Type= 0
Dn Type= 1
Dn Known WS=0.9
Boundary for River Rch & Prof#=Churchill River,Main            , 696
Up Type= 0
Dn Type= 1
Dn Known WS=0.9
Boundary for River Rch & Prof#=Churchill River,Main            , 697
Up Type= 0
Dn Type= 1
Dn Known WS=0.9
Boundary for River Rch & Prof#=Churchill River,Main            , 698
Up Type= 0
Dn Type= 1
Dn Known WS=0.9
Boundary for River Rch & Prof#=Churchill River,Main            , 699
Up Type= 0
Dn Type= 1
Dn Known WS=0.9
Boundary for River Rch & Prof#=Churchill River,Main            , 700
Up Type= 0
Dn Type= 1
Dn Known WS=0.9
Boundary for River Rch & Prof#=Churchill River,Main            , 701
Up Type= 0
Dn Type= 1
Dn Known WS=1
Boundary for River Rch & Prof#=Churchill River,Main            , 702
Up Type= 0
Dn Type= 1
Dn Known WS=1
Boundary for River Rch & Prof#=Churchill River,Main            , 703
Up Type= 0
Dn Type= 1
Dn Known WS=1
Boundary for River Rch & Prof#=Churchill River,Main            , 704
Up Type= 0
Dn Type= 1
Dn Known WS=1
Boundary for River Rch & Prof#=Churchill River,Main            , 705
Up Type= 0
Dn Type= 1
Dn Known WS=1
Boundary for River Rch & Prof#=Churchill River,Main            , 706
Up Type= 0
Dn Type= 1
Dn Known WS=1
Boundary for River Rch & Prof#=Churchill River,Main            , 707
Up Type= 0
Dn Type= 1
Dn Known WS=1
Boundary for River Rch & Prof#=Churchill River,Main            , 708
Up Type= 0
Dn Type= 1
Dn Known WS=1
Boundary for River Rch & Prof#=Churchill River,Main            , 709
Up Type= 0
Dn Type= 1
Dn Known WS=1
Boundary for River Rch & Prof#=Churchill River,Main            , 710
Up Type= 0
Dn Type= 1
Dn Known WS=1
Boundary for River Rch & Prof#=Churchill River,Main            , 711
Up Type= 0
Dn Type= 1
Dn Known WS=1
Boundary for River Rch & Prof#=Churchill River,Main            , 712
Up Type= 0
Dn Type= 1
Dn Known WS=1
Boundary for River Rch & Prof#=Churchill River,Main            , 713
Up Type= 0
Dn Type= 1
Dn Known WS=1
Boundary for River Rch & Prof#=Churchill River,Main            , 714
Up Type= 0
Dn Type= 1
Dn Known WS=1
Boundary for River Rch & Prof#=Churchill River,Main            , 715
Up Type= 0
Dn Type= 1
Dn Known WS=1
Boundary for River Rch & Prof#=Churchill River,Main            , 716
Up Type= 0
Dn Type= 1
Dn Known WS=1
Boundary for River Rch & Prof#=Churchill River,Main            , 717
Up Type= 0
Dn Type= 1
Dn Known WS=1
Boundary for River Rch & Prof#=Churchill River,Main            , 718
Up Type= 0
Dn Type= 1
Dn Known WS=1
Boundary for River Rch & Prof#=Churchill River,Main            , 719
Up Type= 0
Dn Type= 1
Dn Known WS=1
Boundary for River Rch & Prof#=Churchill River,Main            , 720
Up Type= 0
Dn Type= 1
Dn Known WS=1
Boundary for River Rch & Prof#=Churchill River,Main            , 721
Up Type= 0
Dn Type= 1
Dn Known WS=1
Boundary for River Rch & Prof#=Churchill River,Main            , 722
Up Type= 0
Dn Type= 1
Dn Known WS=1
Boundary for River Rch & Prof#=Churchill River,Main            , 723
Up Type= 0
Dn Type= 1
Dn Known WS=1
Boundary for River Rch & Prof#=Churchill River,Main            , 724
Up Type= 0
Dn Type= 1
Dn Known WS=1
Boundary for River Rch & Prof#=Churchill River,Main            , 725
Up Type= 0
Dn Type= 1
Dn Known WS=1
Boundary for River Rch & Prof#=Churchill River,Main            , 726
Up Type= 0
Dn Type= 1
Dn Known WS=1
Boundary for River Rch & Prof#=Churchill River,Main            , 727
Up Type= 0
Dn Type= 1
Dn Known WS=1
Boundary for River Rch & Prof#=Churchill River,Main            , 728
Up Type= 0
Dn Type= 1
Dn Known WS=1
Boundary for River Rch & Prof#=Churchill River,Main            , 729
Up Type= 0
Dn Type= 1
Dn Known WS=1
Boundary for River Rch & Prof#=Churchill River,Main            , 730
Up Type= 0
Dn Type= 1
Dn Known WS=1
Boundary for River Rch & Prof#=Churchill River,Main            , 731
Up Type= 0
Dn Type= 1
Dn Known WS=1
Boundary for River Rch & Prof#=Churchill River,Main            , 732
Up Type= 0
Dn Type= 1
Dn Known WS=1
Boundary for River Rch & Prof#=Churchill River,Main            , 733
Up Type= 0
Dn Type= 1
Dn Known WS=1
Boundary for River Rch & Prof#=Churchill River,Main            , 734
Up Type= 0
Dn Type= 1
Dn Known WS=1
Boundary for River Rch & Prof#=Churchill River,Main            , 735
Up Type= 0
Dn Type= 1
Dn Known WS=1
DSS Import GetInterval= 0
DSS Import GetPeak= 0
DSS Import FillOption= 0
