HEC-RAS study Churchill_Forecasting.prj: ChurchillRiver_Forecasting

--- Churchill_Forecasting.g11 (geometry) --- (continued)

Type RM Length L Ch R = 1 ,15622.24,502.11,500.14,501.46
XS GIS Cut Line= 2
     379896.7436    5906799.3701380146.0105672965904224.39180596
#Sta/Elev= 30
       0     3.4    89.9    3.46  104.88    1.16  184.79    2.83  274.68    1.16
  339.61    4.87  639.26    2.35  761.59    4.64  777.19    -.75  854.15   -1.03
  883.03    -.15     900     2.8    1050     2.8  1071.2     .56 1303.56   -2.38
  1380.4     .79 1483.28    1.29 1698.04    1.41    1728    4.62 1757.97     .73
 1841.84    1.23 2006.04   -3.21 2057.52   -6.38 2168.37   -4.81 2187.98   -2.35
 2287.24    -.12    2310     2.8    2500     2.8 2577.02    6.65 2587.01   13.05
#Mann= 8 ,-1 , 0
       0    .055       0  761.59   .0285       0     900    .035       0
  1071.2   .0285       0 1483.28    .035       0 1841.84   .0285       0
    2310   .0285       0 2587.01    .055       0
Levee=-1,762.29,4.39,0,,,Levee 9,
Bank Sta=761.59,2587.01
XS Rating Curve= 0 ,0
Exp/Cntr(USF)=0.5,0.3
Exp/Cntr=0.3,0.1

Type RM Length L Ch R = 1 ,15122.1 ,308.62,512.16,677.55
XS GIS Cut Line= 2
     380394.3265    5906848.4833380644.0627147735904268.65853826
#Sta/Elev= 30
       0    1.13  199.76    3.57  444.47    2.53  504.39    3.93  519.38    2.12
  589.29    3.13  619.26    5.98  644.23     3.2  729.12    3.21  739.11    4.53
   913.9    3.04  933.55    -.22  961.21    -.68 1100.61   -1.11 1178.85      .6
 1229.26   -1.52 1481.17   -1.37 1506.16    -.38    1520     2.6 1589.05     .77
 1933.31    1.17    2109   -2.82  2341.3    -2.9 2391.73   -5.21 2436.22   -4.89
 2453.74   -2.06 2520.54    2.06 2529.34    7.61 2566.92    7.21 2591.89   12.21
#Mann= 5 ,-1 , 0
       0    .055       0   913.9   .0285       0    1520    .035       0
 1933.31   .0285       0 2529.34    .055       0
Levee=-1,618.54,5.99,0,,,Levee 9,
Bank Sta=913.9,2529.34
XS Rating Curve= 0 ,0
Exp/Cntr(USF)=0.5,0.3
Exp/Cntr=0.3,0.1

Type RM Length L Ch R = 1 ,14609.94,493.61,494.36,496.64
XS GIS Cut Line= 2
     380673.5607    5906880.9974381237.2363106745904397.48940654
#Sta/Elev= 30
       0   10.07    9.99    9.29   19.97    3.07   34.95    1.23  574.25    3.73
  604.21    1.38  624.19    3.94  654.15    2.97  719.07    5.11   848.9     2.5
  893.84    4.02  913.81     7.3  938.78    3.21 1093.58    4.16 1107.27    3.08
 1131.08    -4.8 1157.77   -7.73 1228.28   -1.76 1325.07   -1.96    1395     2.6
  1692.8    1.47    1910     2.6    2030     2.6 2057.09     .55 2123.53   -1.77
 2278.22    -.55 2418.97   -6.88 2491.35   -6.63  2536.7    8.23 2546.68    8.58
#Mann= 7 ,-1 , 0
       0    .055       0 1093.58   .0285       0    1395    .035       0
  1692.8    .035       0    1910    .035       0 2057.09   .0285       0
  2536.7    .055       0
Levee=-1,914.75,7.32,0,,,Levee 9,
Bank Sta=1093.58,2536.7
XS Rating Curve= 0 ,0
Exp/Cntr(USF)=0.5,0.3
Exp/Cntr=0.3,0.1

Type RM Length L Ch R = 1 ,14115.58,502.3,502.01,505.04
XS GIS Cut Line= 2
381171.5856811245906916.59590779381701.5223553145904581.73902776
#Sta/Elev= 30
   54.99    8.78   74.98    3.46  164.96    1.37  219.95    3.01  279.94    1.43
  309.93    3.13  544.88    1.31  719.84    2.73  744.83    4.34   904.8    2.09
 1134.75    3.99 1154.74    1.95 1161.28   -2.87 1243.36    -4.9 1293.14   -2.61
 1303.42     .63    1350     2.5 1639.63    1.58    1720     2.5 1964.56    1.17
    2040     2.5    2150     2.5 2164.96    -.26 2265.42   -2.31 2316.27   -7.28
 2366.56      -9 2407.79   -7.72 2440.92    1.01 2447.58    6.89 2449.21    6.88
#Mann= 9 ,-1 , 0
   54.99    .055       0 1134.75   .0285       0    1350    .035       0
 1639.63   .0285       0    1720    .035       0 1964.56   .0285       0
    2040    .035       0 2164.96    .025       0 2447.58    .055       0
Levee=-1,1110.77,3.98,0,,,Levee 9,
Bank Sta=1134.75,2447.58
XS Rating Curve= 0 ,0
Exp/Cntr(USF)=0.5,0.3
Exp/Cntr=0.3,0.1

Type RM Length L Ch R = 1 ,13613.57,343.57,506.15,654.42
XS GIS Cut Line= 2
     381642.5406    5907109.1877382196.5057057055904668.46351006
#Sta/Elev= 30
       0    9.81       5   10.13   24.98    2.32  319.72    4.44   339.7    1.33
  494.57    2.79  519.54    1.51  584.49    2.52  714.37    1.51 1191.27    2.72
 1202.68   -2.07 1477.47     .79 1765.13    -.96 1917.23     .63 2112.32   -1.86
 2173.55   -1.07 2179.47     .17 2223.55    -.76 2254.31   -4.09 2264.64   -3.26
 2295.33   -5.97 2325.51   -5.56 2348.79   -7.63 2375.13   -7.27 2395.23   -5.32
 2434.35   -6.28 2444.49   -4.92 2459.76     .98 2467.58    7.34  2502.8    7.82
#Mann= 3 , 0 , 0
       0    .055       0 1191.27   .0285       0 2467.58    .055       0
Levee=-1,1176.1,2.87,0,,,Levee 9,
Bank Sta=1191.27,2467.58
XS Rating Curve= 0 ,0
Exp/Cntr(USF)=0.5,0.3
Exp/Cntr=0.3,0.1

Type RM Length L Ch R = 1 ,13107.42,506.78,506.93,512.59
XS GIS Cut Line= 2
     381956.6837    5907185.7673382774.003128878 5904735.0743965
#Sta/Elev= 30
       0    2.44   19.99    1.75   479.7    3.13  624.61    1.39  779.52    2.81
  894.44    2.03 1069.33    2.86 1084.16    -.08 1273.51   -1.81 1325.72    -.61
    1350     2.4    1470     2.4 1494.07       1    1800     2.4 1829.23    -.12
 1846.97   -1.01 1985.46   -1.03 2015.23     .21    2030     2.4    2120     2.4
 2139.19      .2 2219.94   -5.03 2249.62   -5.63 2320.98   -5.17 2361.43   -3.12
 2492.91   -3.79 2525.24    -.59 2533.97    3.81 2548.41    7.89 2583.39    8.22
#Mann= 7 ,-1 , 0
       0    .055       0 1069.33   .0285       0    1350    .035       0
 1829.23   .0285       0    2030    .035       0 2139.19   .0285       0
 2548.41    .055       0
Levee=-1,1062.85,2.85,0,,,Levee 9,
Bank Sta=1069.33,2548.41
XS Rating Curve= 0 ,0
Exp/Cntr(USF)=0.5,0.3
Exp/Cntr=0.3,0.1

Type RM Length L Ch R = 1 ,12600.49,374.32,499.98,635.01
XS GIS Cut Line= 2
     382438.0603    5907344.0193383292.9487421035904780.67768102
#Sta/Elev= 30
       0    1.78  319.66    2.95  329.65     1.5  439.54    2.54  654.31    1.37
  844.11    2.32     954     4.2  978.97    1.83 1009.25    2.11 1018.85   -1.68
 1148.45      .4  1455.7    -.43 1478.45    1.86 1718.56     .45 1758.41   -2.17
 1933.41     .58    1960     2.3    2140     2.3 2151.17     .32 2171.34   -2.16
 2324.57   -3.52 2396.18   -2.25 2486.94   -5.62 2527.74   -4.38 2557.87   -6.04
 2586.54   -3.41 2602.46    3.23 2622.24    3.98 2692.17    2.64 2702.16    4.72
#Mann= 7 ,-1 , 0
       0    .055       0 1009.25   .0285       0 1478.45    .035       0
 1718.56   .0285       0    1960    .035       0 2151.17   .0285       0
 2602.46    .055       0
Levee=-1,953.33,4.17,-1,2623.52,3.97,Levee 9,Levee 11
Bank Sta=1009.25,2602.46
XS Rating Curve= 0 ,0
Exp/Cntr(USF)=0.5,0.3
Exp/Cntr=0.3,0.1

Type RM Length L Ch R = 1 ,12100.51,507.84,506.64,517.95
XS GIS Cut Line= 2
     382766.0584    5907486.1563383882.9724362735904834.38275725
#Sta/Elev= 30
       0    2.12  429.61    3.22  524.53     .98  814.27    2.61  839.24    1.42
 1028.06     .42  1068.1   -1.88 1227.78     .44  1339.1    -.89 1359.59     .85
 1373.84    -.24    1399     2.3    1775     2.3 1786.65   -1.15 1806.19   -4.85
  1865.5   -5.36 1875.11   -2.53 1946.11    -.97 2221.91   -2.81 2282.48    -.39
 2593.96   -4.75  2604.1   -3.33 2624.62   -5.23 2654.18   -4.44 2677.52    3.88
 2732.54    3.16 2752.52    4.32 2847.44     3.1 2862.43    1.52 2877.41    4.77
#Mann= 5 ,-1 , 0
       0    .055       0  814.27   .0285       0    1399    .035       0
 1786.65   .0285       0 2677.52    .055       0
Levee=-1,814.65,2.59,-1,2700.68,4.44,Levee 9,Levee 11
Bank Sta=814.27,2677.52
XS Rating Curve= 0 ,0
Exp/Cntr(USF)=0.5,0.3
Exp/Cntr=0.3,0.1

Type RM Length L Ch R = 1 ,11593.87,500.02,500.21,510.72
XS GIS Cut Line= 2
 383237.132849855907671.67422207384538.3860898175904582.24324925
#Sta/Elev= 30
   24.98    7.97   39.97    1.51  144.88    2.89  184.85    1.23  449.63    2.53
  459.63     .85  519.58    2.25  649.47    1.47  764.38     2.8   859.3    1.56
 1233.97    1.72 1308.37   -3.75 1398.27   -2.13 1438.68     .54 1467.52    -.42
 1498.12   -4.11 1618.06   -4.67 1696.26     .06 1918.41     .51    1935     2.2
    2150     2.2 2166.39     .48 2408.88    -.33 2499.89   -2.82 2661.77   -3.54
 2694.65   -2.41 2716.07    2.78  3072.5    3.85 3362.26    2.57 3377.25    4.89
#Mann= 5 ,-1 , 0
   24.98    .055       0 1233.97   .0285       0    1935    .035       0
 2166.39   .0285       0 2716.07    .055       0
Levee=-1,1209.75,2.42,-1,2742.75,3.17,Levee 9,Levee 11
#XS Ineff= 2 , 0
         1208.84    2.45
Permanent Ineff=
       F       F
Bank Sta=764.38,2716.07
XS Rating Curve= 0 ,0
Exp/Cntr(USF)=0.5,0.3
Exp/Cntr=0.3,0.1

Type RM Length L Ch R = 1 ,11093.66,491.8,491.97,502.32
XS GIS Cut Line= 2
383807.9580584745907604.52322911385032.3599334045904697.55254782
#Sta/Elev= 30
  319.93    8.79  339.93    1.34  589.87    2.02  659.85     .96  679.85    2.74
  829.82    1.91  883.79    2.86     900       2 1182.45    1.28 1245.39   -2.47
 1307.02    -.79 1357.95   -2.84 1439.62   -2.94 1694.85   -1.69 1755.94     .79
  1816.3    -.91 1997.19    -.04    2020       2    2305       2 2345.31     .51
 2466.34   -2.22 2547.56   -1.64 2703.86   -4.18 2732.63    -3.7 2751.84    3.09
 3009.34    3.29 3064.32    1.88 3099.31    4.04 3449.24    2.59 3474.23    7.05
#Mann= 7 ,-1 , 0
  319.93    .055       0  883.79   .0285       0     900    .035       0
 1182.45   .0285       0    2020    .035       0 2345.31   .0285       0
 2751.84    .055       0
Levee=-1,787.18,3.03,-1,2949.6,3.73,Levee 9,Levee 11
Bank Sta=883.79,2751.84
XS Rating Curve= 0 ,0
Exp/Cntr(USF)=0.5,0.3
Exp/Cntr=0.3,0.1

Type RM Length L Ch R = 1 ,10601.69,526.02,523.72,530.89
XS GIS Cut Line= 2
384301.0055540255907700.86502134385465.0994229265904937.07748273
#Sta/Elev= 30
  429.85     7.7  444.84    3.42  484.83    5.66  509.82    5.11  544.81    6.14
  689.76    5.28  798.93    3.87 1299.47   -3.14 1350.44   -2.71 1422.37     -.1
 1552.04   -1.89 1622.46    -1.7 1682.26    -.09    1710       2    2470       2
 2488.12     .75 2498.41   -2.17  2508.4   -3.12 2559.13   -4.08  2689.2    -1.8
 2780.11   -2.44 2804.01    3.05 3098.91    2.81 3168.89    3.62 3178.88    4.62
 3273.85    2.91 3328.83     3.7  3413.8    2.42  3418.8    5.56  3428.8    6.79
#Mann= 5 ,-1 , 0
  429.85    .055       0  798.93   .0285       0    1710    .035       0
 2488.12   .0285       0 2804.01    .055       0
Levee=-1,575.61,5.93,-1,3186.06,4.74,Levee 9,Levee 11
Bank Sta=689.76,2804.01
XS Rating Curve= 0 ,0
Exp/Cntr(USF)=0.5,0.3
Exp/Cntr=0.3,0.1

Type RM Length L Ch R = 1 ,10077.97,521.17,511.58,513.31
XS GIS Cut Line= 2
384898.0292449925907629.68823968 385917.752832965905208.66400365
#Sta/Elev= 30
  739.16     6.1  784.11     5.7  804.09    5.31  814.08    2.64  826.78   -4.24
  927.22    -.59 1105.96   -3.14 1145.18   -2.27 1168.67    1.81 1283.54    2.08
 1354.91     .04 1569.39   -1.65 1768.62     .18 1828.84   -2.69 1849.01   -2.59
 1868.77    -.35 1928.43   -1.28    1990     1.7    2340     1.7 2370.21   -1.01
 2509.08     .52 2900.01   -2.77 2936.67    3.18 3101.48    3.07  3176.4    1.39
 3211.36    3.17 3256.31    1.52 3336.22    3.23 3346.21    5.41 3366.18    6.52
#Mann= 7 ,-1 , 0
  739.16    .055       0  784.11   .0285       0 1168.67    .035       0
 1283.54   .0285       0    1990    .035       0 2370.21   .0285       0
 2936.67    .055       0
Levee=0,,,-1,2986.93,3.24,,Levee 11
Bank Sta=804.09,2936.67
XS Rating Curve= 0 ,0
Exp/Cntr(USF)=0.5,0.3
Exp/Cntr=0.3,0.1

Type RM Length L Ch R = 1 ,9566.389,526.44,517.03,518.5
XS GIS Cut Line= 2
385449.7997380945907631.53848298386524.0371976565905081.08760957
#Sta/Elev= 30
 1029.06    6.28 1084.01    5.64 1098.99    2.08 1109.18    -3.2 1119.08   -6.25
 1243.67   -1.12 1284.32   -1.36 1327.92     .58 1373.74    2.23 1403.71     .13
  1413.7    1.58 1488.64    2.28 1498.63     .55 1574.67    -.22 1886.65   -1.04
 1938.64   -4.26 1976.05   -4.63 2007.33    -1.1 2027.41    -.24 2127.86    -.06
    2140     1.5    2820     1.5 2837.14     .65 2937.68   -1.03 2957.71   -3.23
 3022.05   -4.32 3066.55   -2.12 3098.76    2.12 3631.68    6.05 3796.52     6.3
#Mann= 7 ,-1 , 0
 1029.06    .055       0 1084.01    .025       0 1327.92    .035       0
 1574.67    .025       0    2140    .035       0 2837.14    .025       0
 3098.76     .05       0
Levee=-1,992.53,6.21,-1,3649.66,6.06,Levee 12,Levee 11
Bank Sta=1084.01,3098.76
XS Rating Curve= 0 ,0
Exp/Cntr(USF)=0.5,0.3
Exp/Cntr=0.3,0.1

Type RM Length L Ch R = 1 ,9049.357,354.9,499.13,661.51
XS GIS Cut Line= 2
 385939.925172245907792.99225504 386897.77358476 5905518.8719472
#Sta/Elev= 30
 1188.85    5.37 1248.79     3.6 1258.78    4.35 1303.36   -1.99 1416.97    -3.3
 1456.65   -4.93 1486.76   -7.45 1517.45    -.96 1709.48   -1.78  1872.4    -.39
 2176.28   -1.89 2216.36    -.51 2236.34   -1.75    2250     1.1    2960     1.1
 2984.65   -1.44 3196.95    -.72 3248.71   -3.38 3279.04   -3.03 3301.79    3.19
 3306.79    3.32 3341.76     2.3  3401.7    2.42 3411.69    1.49 3426.67    2.02
 3436.66     .89 3506.59    2.89 3616.49    2.11 3631.47    5.15 3656.45    5.56
#Mann= 5 ,-1 , 0
 1188.85    .055       0 1258.78    .025       0    2250    .035       0
 2984.65    .025       0 3306.79     .05       0
Levee=0,,,-1,3304.29,3.14,,Levee 11
Bank Sta=1258.78,3301.79
XS Rating Curve= 0 ,0
Exp/Cntr(USF)=0.5,0.3
Exp/Cntr=0.3,0.1

Type RM Length L Ch R = 1 ,8550.231,401.22,484.88,570.88
XS GIS Cut Line= 2
 386223.317029655908162.16379178387469.8446558355905717.89075788
#Sta/Elev= 30
 1034.53   10.72  1094.5   10.18  1099.5    9.75 1124.65    -.96    1160      .4
 1275.53     .21 1443.08   -5.01 1563.68   -2.93    1600     1.1    2060     1.1
 2078.92    -.18 2299.18   -2.51 2330.35   -1.76    2350     1.7 3163.57     .83
 3193.56    2.83 3223.54    1.28 3238.54    2.53 3318.57    1.83 3331.32    -.74
 3336.26   -2.09 3364.92   -3.12 3513.83   -2.23  3527.3    1.78  3548.4    1.85
 3648.35    2.87 3713.32     .46 3748.31    2.26 3753.31    4.58  3778.3    5.68
#Mann= 7 ,-1 , 0
 1034.53    .055       0  1094.5    .025       0    1600    .035       0
 2078.92    .025       0    2350    .035       0 3331.32    .025       0
  3548.4     .05       0
Bank Sta=1094.5,3527.3
XS Rating Curve= 0 ,0
Exp/Cntr(USF)=0.5,0.3
Exp/Cntr=0.3,0.1

Type RM Length L Ch R = 1 ,8065.351,440.96,519.76,595.84
XS GIS Cut Line= 2
386562.6949334715908436.15059991387968.2569076065905928.98040802
#Sta/Elev= 30
  994.76    9.44 1018.68    -1.5 1028.28   -3.74 1055.78   -2.08 1065.55    -.25
 1100.71    -.01 1156.31   -3.87 1207.61   -1.67 1300.48    -.26 1475.35   -1.98
 1762.15   -1.83 1801.06   -5.13 1831.54   -1.08 2031.91   -1.66 2271.35    .002
    2290     1.1    3050     1.1 3104.25     1.3 3114.25    2.16 3169.23     2.5
 3214.22     1.4  3294.2    2.66 3469.16    1.01 3534.14    2.41 3587.32   -1.15
 3638.18   -2.05 3790.57   -2.01 3828.24   -1.13 3864.06    4.23 3869.06    4.33
#Mann= 5 ,-1 , 0
  994.76     .02       0    2290    .035       0 3114.25    .035       0
 3587.32    .025       0 3864.06     .05       0
Bank Sta=994.76,3864.06
XS Rating Curve= 0 ,0
Exp/Cntr(USF)=0.5,0.3
Exp/Cntr=0.3,0.1

Type RM Length L Ch R = 1 ,7545.588,500.9,504.07,503.17
XS GIS Cut Line= 2
386910.6886386165908760.28079192388532.2559101445906085.77140968
#Sta/Elev= 30
  929.32    7.94  939.31    7.65  952.29    1.75  971.85   -2.74 1001.24   -2.76
    1020     1.1    1610     1.1 1622.14     -.2 1771.09   -1.41 1777.66   -3.04
 1821.25    -3.6 1871.01   -6.33 1911.96   -6.21 1973.58   -3.47 1993.86    -.44
 2084.04    -.26    2110     1.1 3417.49    1.61 3430.48   -1.12 3462.45   -2.64
 3564.48   -2.27 3579.49    2.71 3902.13    1.92 3925.84    -4.5 3980.98   -2.45
 3997.06    1.68 4022.05    1.06 4032.04    3.54 4052.02    4.64 4057.02    4.96
#Mann= 9 ,-1 , 0
  929.32    .055       0  939.31    .025       0    1020    .035       0
 1622.14    .025       0    2110    .035       0 3417.49    .025       0
 3579.49    .035       0 3925.84    .025       0 4052.02     .05       0
Bank Sta=939.31,4052.02
XS Rating Curve= 0 ,0
Exp/Cntr(USF)=0.5,0.3
Exp/Cntr=0.3,0.1

Type RM Length L Ch R = 1 ,7041.521,669.66,508.05,362.61
XS GIS Cut Line= 2
387268.1470556665909134.01635898389096.9485152045906117.70818616
#Sta/Elev= 30
   819.4    9.83  834.39    8.99  858.12   -2.09     940     1.1    1184     1.1
  1204.9   -1.26 1488.89    -.93 1508.96   -2.48 1675.45    -.58  2083.3   -3.52
 2113.31   -1.44 2402.29    -.45 2705.27   -2.65 2939.28    -.55 3058.58   -1.81
 3069.58       1  3075.1    4.54    3100     1.1    3300     1.1 3333.08   -2.17
 3452.88   -1.01 3502.45    1.92  3562.4     3.1 3747.27    1.42 4052.05    1.73
 4068.84   -1.88 4117.36   -4.18  4130.8   -2.84 4140.89    3.73 4346.84    4.23
#Mann= 9 ,-1 , 0
   819.4    .055       0  834.39    .025       0     940    .035       0
  1204.9    .025       0 3069.58    .035       0 3333.08    .025       0
 3502.45    .035       0 4068.84    .025       0 4140.89     .05       0
Bank Sta=834.39,4140.89
XS Rating Curve= 0 ,0
Exp/Cntr(USF)=0.5,0.3
Exp/Cntr=0.3,0.1

Type RM Length L Ch R = 1 ,6533.468,735.32,475.47,238.27
XS GIS Cut Line= 2
387805.7468626965909456.11270313389352.748295061 5906476.7372939
#Sta/Elev= 30
  799.33    9.79 1261.04    -.23 1308.95   -2.06 1348.12   -4.42 1377.09   -4.26
 1387.38   -1.62 1415.61   -1.07 1482.83   -3.79 1613.31    -1.3 1968.46   -1.76
  1998.8   -1.19    2020     1.1    3070     1.1 3090.27     .09 3138.69   -1.74
 3167.99   -1.84 3226.33    -.35 3297.14    -.93 3306.89    -2.3 3369.07   -2.83
 3402.04    1.42  3686.8    1.62 3721.77    1.43 3731.76     .38 3756.73    1.68
 3976.54    2.03 3992.85   -2.55 4052.16   -3.97 4081.45    3.64 4156.39    4.06
#Mann= 6 ,-1 , 0
  799.33     .02       0    2020    .035       0 3090.27    .025       0
 3402.04    .035       0 3992.85    .025       0 4081.45     .05       0
Bank Sta=799.33,4081.45
XS Rating Curve= 0 ,0
Exp/Cntr(USF)=0.5,0.3
Exp/Cntr=0.3,0.1

Type RM Length L Ch R = 1 ,6057.999,902.53,464.84,160.09
XS GIS Cut Line= 2
388461.2716433575909637.87214471389588.5124833875906724.74443417
#Sta/Elev= 30
  919.58    9.21 1017.16   -2.23    1160      .6    1350      .6 1378.03   -1.82
 1526.29   -3.37 1557.22    -7.3  1567.4    -4.7 1587.69   -6.16 1618.16   -5.42
 1638.63   -3.31 1734.21    1.15    2235      .6    3000      .6 3003.22    -.54
 3067.45    -.93    3087      .6    3423      .6 3453.43    1.86 3588.37     .67
 3643.35    1.12 3653.34    2.41 3853.26       0 3883.24    1.68 3933.22    1.72
 3951.43   -3.52 3986.95   -3.08  4003.3     .22 4008.27    3.25 4043.17    3.55
#Mann= 10 ,-1 , 0
  919.58     .02       0    1160    .035       0 1378.03    .025       0
 1734.21    .035       0    2235    .035       0 3003.22    .025       0
    3087    .035       0 3453.43    .035       0 3933.22    .025       0
 4008.27     .05       0
Bank Sta=919.58,4008.27
XS Rating Curve= 0 ,0
Exp/Cntr(USF)=0.5,0.3
Exp/Cntr=0.3,0.1

Type RM Length L Ch R = 1 ,5593.158,526.82,512.81,384.54
XS GIS Cut Line= 2
389250.1617883315909671.42304574 389755.785370025906807.62898116
#Sta/Elev= 30
 1138.77    7.82 1141.74    7.57 1153.27     .04 1167.07   -3.33 1197.04   -1.64
 1317.54    -.44 1337.52   -3.48 1511.71   -4.13 1753.84   -2.17 1794.09   -1.11
 1822.49    1.86 2012.44    1.19  2035.9   -2.06 2051.49   -2.44    2150       1
    2859       1  2879.7   -1.16    2905    -.33 3012.18   -1.85    3032       1
 3741.94    1.25 3765.71   -2.76 3823.92   -3.18 3861.54   -2.33 3897.37   -3.45
 3907.15   -1.84 3921.11   -3.51 3931.72     .41 3931.72     3.6 4046.85    3.85
#Mann= 8 ,-1 , 0
 1138.77     .02       0 1822.49    .035       0 2012.44    .025       0
    2150    .035       0  2879.7    .025       0    3032    .035       0
 3741.94    .025       0 3931.72     .05       0
Bank Sta=1141.74,3931.72
XS Rating Curve= 0 ,0
Exp/Cntr(USF)=0.5,0.3
Exp/Cntr=0.3,0.1

Type RM Length L Ch R = 1 ,5080.352,171.62,526.28,896.9
XS GIS Cut Line= 2
389773.3241114275909556.74655967390190.7926560965907159.37884481
#Sta/Elev= 30
 1414.09    7.32 1424.08    7.08 1434.07    2.35 1444.07    1.12 1474.05    2.36
 1489.04    1.01 1509.03    1.69 1518.22   -4.55 1528.07   -7.17 1533.68  -11.38
 1544.53  -11.24 1611.14   -2.94 1851.16    -.14 1860.67    -.94    1880      .8
    2853      .8 2873.86   -1.11 3044.15   -3.08 3155.87    -.93 3242.44   -2.18
 3326.62    -.39    3491   -1.69    3515      .8    3690      .8  3719.2    -1.4
 3736.51   -1.79 3767.56    2.04 3777.56     .96 3792.55    3.75 3847.51    3.97
#Mann= 7 ,-1 , 0
 1414.09    .055       0 1424.08    .025       0    1880    .035       0
 2873.86    .025       0    3515    .035       0  3719.2    .025       0
 3792.55     .05       0
Bank Sta=1424.08,3792.55
XS Rating Curve= 0 ,0
Exp/Cntr(USF)=0.5,0.3
Exp/Cntr=0.3,0.1

Type RM Length L Ch R = 1 ,4554.075,342.12,461.93,591.45
XS GIS Cut Line= 2
390028.8622690035909883.80463814390793.2241185295907625.73349269
#Sta/Elev= 30
 1164.47    7.11 1174.47     6.8 1179.47    6.78 1192.64   -7.31 1204.46    -9.7
    1262   -2.13 1270.28      -4 1310.23   -5.81 1386.11   -7.73 1464.99   -5.84
 1473.59   -8.28 1520.19   -4.96  1534.3     1.6 1689.24    2.16 1704.87   -5.39
 1724.43   -8.17 1803.21   -7.55 1851.89   -1.41 2284.66   -1.13 2314.93   -2.38
 2436.28   -1.87    2456      .8    3118      .8 3138.88    -.94 3367.75   -3.14
 3396.49    -.77 3507.35     .01 3510.28    1.59  3538.4    2.11 3548.39    4.03
#Mann= 7 ,-1 , 0
 1164.47    .055       0 1174.47    .025       0  1534.3    .035       0
 1689.24    .025       0    2456    .035       0 3138.88    .025       0
 3548.39     .05       0
Bank Sta=1179.47,3548.39
XS Rating Curve= 0 ,0
Exp/Cntr(USF)=0.5,0.3
Exp/Cntr=0.3,0.1

Type RM Length L Ch R = 1 ,4092.149,230.75,459.45,666.47
XS GIS Cut Line= 2
390376.2427330745910066.05904151391225.2543586975907941.08811592
#Sta/Elev= 30
 1169.12    5.75 1184.11     .91  1204.1    1.26 1236.84     .44 1276.37   -6.58
 1334.73   -6.11 1354.81   -1.19 1364.47   -2.35 1401.23   -1.38 1423.93    1.54
 1628.78    1.37 1643.77     .06 1673.75    3.96 1713.72    1.34 1803.41    1.99
 1807.73      .7 1928.77      -3 2111.08   -3.78 2181.66   -9.67 2200.76   -3.21
 2359.12   -1.52    2380      .8 2904.74      .6 2960.81   -2.88 3307.09   -1.72
 3348.38    -8.7 3358.62   -8.81 3391.84    -.04 3398.77    5.52 3457.41    6.15
#Mann= 7 ,-1 , 0
 1169.12    .055       0  1204.1    .025       0 1423.93    .035       0
 1803.41    .025       0    2380    .035       0 2904.74    .025       0
 3398.77     .05       0
Bank Sta=1204.1,3398.77
XS Rating Curve= 0 ,0
Exp/Cntr(USF)=0.5,0.3
Exp/Cntr=0.3,0.1

Type RM Length L Ch R = 1 ,3632.701,300.31,466.67,610.79
XS GIS Cut Line= 2
390636.7859122825910279.42911882391933.7067771495907812.47081517
#Sta/Elev= 30
 1118.83     4.9  1148.8    3.85 1158.79     1.4 1268.67    1.31 1299.91   -4.11
  1330.2   -3.22 1398.96   -6.57 1418.39    -.37  1430.3     .66 1798.12     .46
 1828.09    2.21 1863.05     .42    2120      .8 2139.16   -1.73    2641   -4.32
 2733.99   -7.09 2756.27   -6.49    2795      .8    3100      .8 3124.71   -1.44
 3236.67    -.83 3287.74   -4.59 3466.35   -3.65 3489.02   -3.03 3507.02    2.53
 3526.31    3.15 3746.08    1.04 3761.06    3.24 3885.93    2.87 3905.91    5.13
#Mann= 7 ,-1 , 0
 1118.83    .055       0 1268.67    .025       0  1430.3    .035       0
 2139.16    .025       0    2795    .035       0 3124.71    .025       0
 3526.31    .055       0
Levee=-1,1120.1,4.85,-1,3525.2,3.08,Levee 13,Levee 14
Bank Sta=1268.67,3507.02
XS Rating Curve= 0 ,0
Exp/Cntr(USF)=0.5,0.3
Exp/Cntr=0.3,0.1

Type RM Length L Ch R = 1 ,3166.035,68.41,461.7,899.38
XS GIS Cut Line= 2
390483.5749218815911210.51167892392442.0912198995908101.93129383
#Sta/Elev= 30
  249.94    4.03  459.89    3.31  514.87    1.86  659.84    2.62  704.83     .07
  759.82    -.17  924.78     2.1 1059.74     1.3 1079.74    2.79 1109.73    -.01
 1149.72    2.19 1184.71     .66  1224.7    1.54  1234.7    1.42 1265.75   -3.73
 1313.75   -4.12 1410.68   -2.32 1424.65    1.49    1670     2.2    1874      .8
 2444.87    -.07 2514.75   -1.19 2714.23    -.87 3067.77    -4.3 3351.57   -3.45
 3427.21   -5.04 3432.73   -2.68 3469.57    1.56 3854.07    1.22 3924.05    3.58
#Mann= 6 ,-1 , 0
  249.94    .055       0  1224.7    .025       0 1424.65    .025       0
    1874    .035       0 2444.87    .025       0 3469.57     .05       0
Levee=-1,1084.74,2.94,0,,,Levee 13,
Bank Sta=1224.7,3469.57
XS Rating Curve= 0 ,0
Exp/Cntr(USF)=0.5,0.3
Exp/Cntr=0.3,0.1

Type RM Length L Ch R = 1 ,2704.339,128.41,458.02,647.53
XS GIS Cut Line= 5
390546.482932983 5911240.2147802      390827.651     5910815.629
     391054.1582    5910597.9076     392772.7882    5908945.9397
392902.1857969325908821.56116645
#Sta/Elev= 30
  264.61    4.09  494.27     -.1  574.15    -.09  614.09    1.91 1028.19    1.09
 1048.14    2.22 1118.02     .28 1197.98    1.34 1241.56   -4.92 1297.72   -5.31
 1321.59    -.44 1323.08     1.2 1629.91     .69    1676      .7  2162.2     .25
    2185      .7    2580      .7 2607.48    -.53 2636.87   -1.51 2881.73    -.85
 2929.38   -2.51 3007.52   -2.56 3038.08   -5.43 3101.79   -6.07 3242.48   -5.88
 3271.66   -4.57 3340.77   -5.44 3380.81   -3.04 3399.84     .95 3651.36    2.71
#Mann= 9 ,-1 , 0
  264.61    .055       0 1197.98    .025       0 1323.08    .035       0
 1629.91    .025       0    1676    .035       0  2162.2    .025       0
    2185    .035       0 2607.48    .025       0 3399.84     .05       0
Levee=-1,1017.42,2.63,0,,,Levee 13,
Bank Sta=1197.98,3399.84
XS Rating Curve= 0 ,0
Exp/Cntr(USF)=0.5,0.3
Exp/Cntr=0.3,0.1

Type RM Length L Ch R = 1 ,2246.315,201.07,447.73,682.36
XS GIS Cut Line= 5
390602.0439653975911386.35436667     390604.7077    5911382.2168
     391119.4203    5910977.8704     393002.1305    5909498.8561
393064.9786581125909449.48402307
#Sta/Elev= 30
  167.25    3.84  207.15    3.33  247.12    -.14  292.09     .12  337.06    2.12
  921.68    1.77  931.68    2.95  966.67    1.07 1044.13    1.55 1060.28   -2.26
 1079.71   -3.58 1146.87   -5.15 1151.37    -.48 1155.11   -3.44 1168.14     1.2
    1415     1.2 1435.84     .18    1460      .6    2635      .6 2655.37    -.67
 2685.18   -2.86 2735.84   -2.18 2786.97   -7.19 2921.46   -5.41 3013.13   -6.52
 3090.88   -5.57  3107.6   -3.25 3146.49   -2.22 3170.91    1.96 3300.82    1.89
#Mann= 7 ,-1 , 0
  167.25    .055       0 1044.13    .025       0 1168.14    .025       0
 1435.84    .025       0    1460    .035       0 2655.37    .025       0
 3170.91     .05       0
Levee=-1,936.53,2.93,-1,3182.95,2,Levee 13,Levee 15
Bank Sta=1044.13,3170.91
XS Rating Curve= 0 ,0
Exp/Cntr(USF)=0.5,0.3
Exp/Cntr=0.3,0.1

Type RM Length L Ch R = 1 ,1798.588,304.53,463.59,618.77
XS GIS Cut Line= 2
390637.0621078185911589.11775628393271.2730150155910017.30875395
#Sta/Elev= 30
   19.98    3.53   54.96    -.07   64.95    2.19  114.91     .08  219.82    2.01
  434.65    1.17  444.64     .23  474.61    1.32  819.34    2.21  924.25     .35
  959.22    1.56 1079.12    1.05 1090.51   -3.66 1100.51   -3.17 1110.43   -6.96
 1182.54   -3.02 1263.96   -1.73 1278.38     .33    1310      .6    2485      .6
 2498.16    -.59 2535.72     -.9 2545.77   -4.43 2565.72   -5.97 2718.78   -6.34
 2810.65   -4.93 2952.61    -7.1  2981.6    -.11 2987.67    2.78  3087.5    3.36
#Mann= 5 ,-1 , 0
   19.98    .055       0 1079.12    .025       0    1310    .035       0
 2498.16    .025       0 2987.67     .05       0
Levee=-1,896.08,2.13,0,,,Levee 13,
Bank Sta=1079.12,2987.67
XS Rating Curve= 0 ,0
Exp/Cntr(USF)=0.5,0.3
Exp/Cntr=0.3,0.1

Type RM Length L Ch R = 1 ,1334.995,253.1,460.22,659.21
XS GIS Cut Line= 2
 390792.220074915911834.79118767393465.0882618155910531.40471842
#Sta/Elev= 30
   64.97    4.07   99.96    -.08  219.91    2.13  479.79    1.92  484.79     .39
  814.65     .92  844.64    2.27 1271.83     .81 1304.79   -2.65 1456.24   -1.33
    1490      .5    1550      .5 1572.79    -1.3 1899.07    -.83 2106.24   -2.97
 2125.52    -1.5 2154.84    -4.1 2174.77   -1.37 2248.47   -1.12 2312.62   -3.89
 2419.44   -4.48 2488.46   -2.79 2718.44   -4.24 2771.74   -7.79 2842.63   -8.43
 2862.62    -5.3 2891.47   -7.16 2939.42    -.21 2945.11    1.88 3038.69     2.3
#Mann= 5 ,-1 , 0
   64.97    .055       0 1271.83    .025       0    1490    .035       0
 1572.79    .025       0 2945.11     .05       0
Levee=-1,886.75,2.21,0,,,Levee 13,
Bank Sta=1271.83,2945.11
XS Rating Curve= 0 ,0
Exp/Cntr(USF)=0.5,0.3
Exp/Cntr=0.3,0.1

Type RM Length L Ch R = 1 ,874.7763,130.1,392.59,756.18
XS GIS Cut Line= 2
390945.7688758475912033.34841432393889.1190668035910970.79641399
#Sta/Elev= 30
  169.96    4.03  259.94    -.09  314.93     -.1  329.92     1.7   439.9     .17
  504.88    1.95 1014.76     .33 1054.75    1.72 1443.96    2.58 1456.32    -.79
 1485.34    -.28 1539.55   -2.71 1723.42    -.89 1813.77    -.86  1863.6   -2.51
 1894.03    -.71 1977.21   -2.28 2037.84   -1.52 2057.93   -5.59 2186.72   -6.73
 2206.94   -4.24 2226.61   -5.57 2246.48   -3.66 2355.05   -6.12 2503.01   -6.66
 2914.17    -.31 2954.33   -1.37 3005.48    -.18 3020.78    1.57 3299.23    4.99
#Mann= 3 , 0 , 0
  169.96     .05       0 1443.96    .025       0 3020.78     .05       0
Levee=-1,1387.68,3.02,0,,,Levee 13,
Bank Sta=1443.96,3020.78
XS Rating Curve= 0 ,0
Exp/Cntr(USF)=0.5,0.3
Exp/Cntr=0.3,0.1

Type RM Length L Ch R = 1 ,482.1884,112.67,449.24,772.32
XS GIS Cut Line= 6
390873.5266551075912193.57600555      391553.291    5911960.6071
     392048.4026     5911878.808     392049.5722    5911878.6148
     393653.9463    5911613.5507393658.868451062 5911612.7374948
#Sta/Elev= 30
   54.89    4.63  139.72    3.64  169.66    1.75  264.48    1.82  369.27     .08
  409.19    1.14  444.12     .15   454.1    1.57  499.01     .25  648.71    1.38
   708.6     .28  723.57    1.77  897.68    1.81  927.49     .75  962.27    1.99
 1406.43    1.38 1433.33     -.5 1846.32   -2.06 1866.93   -6.79  1959.3    -8.8
 2021.33   -6.01 2226.43   -3.67 2297.97   -5.37 2349.14   -3.87 2648.16   -2.42
 2698.07    -.51 2707.23    3.67 2728.01    5.15 2867.68    5.43 2907.59    7.49
#Mann= 3 , 0 , 0
   54.89     .05       0 1406.43    .025       0 2707.23     .05       0
Bank Sta=1406.43,2707.23
XS Rating Curve= 0 ,0
Exp/Cntr(USF)=0.5,0.3
Exp/Cntr=0.3,0.1

Type RM Length L Ch R = 1 ,32.94778,413.74,478.28,640.54
XS GIS Cut Line= 4
     390848.0599    5912303.9762     391122.9355    5912226.9858
     392022.9791    5912202.7855393370.1307005935912166.56340159
#Sta/Elev= 30
       0    4.04  132.88    3.19  260.85      .8  330.22    1.29  350.12     .26
  374.99    1.21  424.74    -.22  454.58    1.38  653.56     .91  683.41    2.48
  907.26     .78  942.08    1.87 1295.63    2.02 1304.89    -.28 1328.88    -.73
 1373.84   -4.75 1391.75    -3.8 1420.65   -6.17 1497.82   -4.55 1527.11   -5.94
 1537.09   -4.21 1566.68   -4.24 1606.47   -6.36 1776.63   -8.54 2212.53    -.39
 2252.57   -1.89 2492.79   -2.76  2517.1     .29 2523.36    4.32 2533.43    4.31
#Mann= 3 , 0 , 0
       0     .06       0 1295.63    .025       0 2523.36     .06       0
Levee=-1,1229,2.12,0,,,Levee 16,
Bank Sta=1295.63,2523.36
XS Rating Curve= 0 ,0
Exp/Cntr(USF)=0.5,0.3
Exp/Cntr=0.3,0.1

Type RM Length L Ch R = 1 ,-445.332,503.69,506.76,490.08
XS GIS Cut Line= 2
     390922.1354    5912619.2117     395604.1073    5912717.8173
#Sta/Elev= 30
       0    3.23  338.46     .69  383.32    1.61  568.12     .44  598.02    1.91
  635.23     .89  672.78    1.63  1140.3    1.49 1175.05  -10.13 1215.24  -10.99
 1235.39   -7.42 1255.77   -5.75 1338.17   -7.19 1511.34   -7.61 1552.43    -4.3
 1702.69    -1.9    1720      .1    2125      .1 2144.61   -1.71 2211.82   -4.23
 2262.08   -4.76 2359.67   -1.98  2518.8    -.94 2668.69   -1.65 2678.72    -.83
    2700     1.5  4063.6     .37 4208.51     1.3 4578.46      .5 4683.01    9.21
#Mann= 5 ,-1 , 0
       0     .06       0  1140.3     .03       0    1720    .045       0
 2144.61     .03       0 2678.72     .06       0
Levee=-1,594.28,1.9,-1,3167.39,1.69,Levee 16,Levee 17
#XS Ineff= 2 , 0
                         3178.96            1.93
Permanent Ineff=
       F       F
Bank Sta=1140.3,2700
XS Rating Curve= 0 ,0
Exp/Cntr(USF)=0.5,0.3
Exp/Cntr=0.3,0.1

Type RM Length L Ch R = 1 ,-952.091,534.3,533.97,511.38
XS GIS Cut Line= 2
     391024.7287    5913099.8707     395599.7588    5913196.2241
#Sta/Elev= 30
       0    2.09   94.92     1.6  104.91     .21  314.73    1.77  454.61    -.19
  609.47    1.77  634.45     .37  799.31    1.48  844.27    -.23   924.2    1.13
 1059.09     .85  1094.3  -10.87 1113.27  -13.15 1123.35  -10.03 1144.23  -14.15
 1194.17   -6.83 1386.91    -3.4    1440      .1    1620      .1  1641.3   -2.37
 1866.78   -2.19    1886      .1    2353      .1 2373.55   -1.43 2510.54   -5.49
 2540.43   -4.81 2572.78    1.02 3891.62    1.08 3961.56    -.34 4576.02    -.32
#Mann= 7 ,-1 , 0
       0    .055       0 1059.09     .03       0    1440    .045       0
  1641.3     .03       0    1886    .045       0 2373.55     .03       0
 2572.78    .055       0
Levee=-1,942.75,1.5,-1,2629.12,1.05,Levee 16,Levee 17
#XS Ineff= 2 , 0
          952.08    1.72 2638.65            1.66
Permanent Ineff=
       F       F
Bank Sta=1059.09,2572.78
XS Rating Curve= 0 ,0
Exp/Cntr(USF)=0.5,0.3
Exp/Cntr=0.3,0.1

Type RM Length L Ch R = 1 ,-1486.06,487.84,486.02,490.18
XS GIS Cut Line= 2
     391133.8455    5913604.0628     395556.5846    5913697.2088
#Sta/Elev= 30
       0    1.87  164.95    2.44  184.95     .96  254.93    1.86  409.88    -.02
  434.87    2.19  459.87     -.4  529.85    1.79  564.84     .65 1148.59    1.09
 1164.66     .72 1191.67   -10.1 1226.86  -11.67  1481.2   -2.19 2112.22   -1.19
 2224.21   -2.28 2264.84   -4.93  2373.8    -5.8 2413.96   -1.57 2645.68   -4.23
 2689.22     .03 2754.21    1.47 2809.19    -.06 2824.19    1.47 2979.14    -.02
 3399.02    1.23 3858.88     .92 3868.88    -.24 4028.83    1.16 4423.72    -.19
#Mann= 3 , 0 , 0
       0     .06       0 1148.59     .03       0 2754.21     .06       0
Levee=-1,1126.32,1.51,-1,2752.21,1.55,Levee 16,Levee 17
#XS Ineff= 2 , 0
         1119.17    1.64 2755.86            1.71
Permanent Ineff=
       F       F
Bank Sta=1148.59,2754.21
XS Rating Curve= 0 ,0
Exp/Cntr(USF)=0.5,0.3
Exp/Cntr=0.3,0.1

Type RM Length L Ch R = 1 ,-1972.08,12000,12000,12000
XS GIS Cut Line= 2
      391501.249    5914089.8532     395361.2289    5914171.1471
#Sta/Elev= 30
       0    1.34  564.39     .98  614.34    -.23  659.29    1.51  719.22     .31
   834.1     .93  889.04    -.33  998.92    -.15 1043.56   -4.29 1157.89   -5.13
  1409.3    -3.6 1611.97   -4.62  1783.5   -2.72 1834.26   -3.33 1864.56   -5.26
 2002.15   -4.63 2040.17    -3.3 2132.08   -7.21 2266.23   -5.03 2367.45    -.16
 3126.63    -.07 3136.62    1.08 3171.58    -.15 3296.45    1.76 3311.43     .56
 3361.38      .5 3381.36     1.6 3456.28     .44 3720.99      .3 3860.84    7.07
#Mann= 3 , 0 , 0
       0     .06       0  998.92     .03       0 2367.45     .06       0
Levee=-1,835.16,0.88,-1,3137.07,1.19,Levee 16,Levee 17
#XS Ineff= 2 , 0
         1009.87     .26 2358.68             .26
Permanent Ineff=
       F       F
Bank Sta=998.92,2367.45
XS Rating Curve= 0 ,0
Exp/Cntr(USF)=0.5,0.3
Exp/Cntr=0.3,0.1

Type RM Length L Ch R = 1 ,-12000  ,0,0,0
XS GIS Cut Line= 5
401323.5326386675923078.93330051401323.5326386675923078.93330051
 402705.653043435920992.72874756404087.7734481925918906.52419462
404087.7734481925918906.52419462
#Sta/Elev= 4
       0       5       5      -5    5000      -5    5005       5
#Mann= 3 , 0 , 0
       0     .06       0       0     .03       0    5005     .06       0
Bank Sta=0,5005
XS Rating Curve= 0 ,0
Exp/Cntr=0.3,0.1

Chan Stop Cuts=-1
Use User Specified Reach Order=0
Composite Channel Slope=5

--- Churchill_Forecasting.g14 (geometry) ---

Geom Title=Current Conditions - Nalcor LiDAR Clip
Program Version=4.10

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
River Reach=Churchill River ,Main

Type RM Length L Ch R = 1 ,41243.44,1199.65,1001.34,790.16
XS GIS Cut Line= 2
355538.233438958 5903210.9299795355305.4634303595900327.36277047
#Sta/Elev= 30
  969.32   24.28  991.86    4.99 1173.44  -21.58 1224.59  -22.69 1265.67  -28.19
 1306.91  -39.04 1376.88  -44.51 1518.59  -44.84  1589.1  -52.43 1659.56  -52.78
 1759.43  -61.63 1891.64  -51.51 1982.31  -35.92 2012.73  -40.16 2063.54  -33.53
 2114.18   -4.89  2287.7     -.7 2357.95   -6.16 2643.14   13.25 2778.97   -9.84
 2799.18  -28.77 2819.15  -36.36 2859.64  -40.41  2971.5  -29.99 3225.62  -23.61
 3407.01   -7.17 3536.99   -5.12 3587.48   12.42 3817.32   18.07 3862.29      29
#Mann= 3 , 0 , 0
  969.32    .055       0  991.86   .0285       0 3587.48    .055       0
Bank Sta=991.86,3587.48
XS Rating Curve= 0 ,0
Exp/Cntr(USF)=0.5,0.3
Exp/Cntr=0.3,0.1

Type RM Length L Ch R = 1 ,39223.7 ,827.11,1029.24,1183.39
XS GIS Cut Line= 2
357556.8319231745902704.63078815357141.5808249635900028.53733652
#Sta/Elev= 30
  914.37   19.11 1104.24   16.75 1164.19    8.79 1174.19    9.85 1189.18   16.08
 1473.98   12.97  1483.5     3.3 1511.85   -1.91 1521.24   -5.75 1612.08   -5.51
 1632.11   -2.62 1662.61   -5.46 1741.73   -4.26 1832.97   -7.52 1873.58   -4.01
  1981.4   -5.56 2123.01   -3.41 2153.71   -6.07 2194.44   -5.99 2378.74   -1.22
 2712.49    1.66 2864.45    1.25 2966.16   -2.26 3219.26      -1 3300.44    1.71
 3410.28     .36 3423.63    3.34 3437.62   14.78 3572.53   15.06 3622.49   20.43
#Mann= 3 , 0 , 0
  914.37    .055       0 1473.98   .0285       0 3437.62    .055       0
Levee=-1,1207.22,16.05,0,,,,
Bank Sta=1473.98,3437.62
XS Rating Curve= 0 ,0
Exp/Cntr(USF)=0.5,0.3
Exp/Cntr=0.3,0.1

Type RM Length L Ch R = 1 ,37189.66,843.23,1008.41,1150.62
XS GIS Cut Line= 2
359179.4351656125901755.21912747359414.2732619825900375.98532351
#Sta/Elev= 30
 1439.07    19.6 1454.06   14.65 1489.04   10.39 1558.99    9.85 1603.96    7.87
 1662.67    8.25 1669.03    3.31 1677.84    2.15 1688.12   -2.64 1809.45    -.44
 2063.59     .07 2174.82   -3.18 2265.79   -2.98 2285.66     .62  2316.4    -.77
 2326.42   -2.84 2366.79   -2.78 2498.76     .65 2559.72    -.66 2641.36    -.29
 2661.18   -1.33 2671.24   -3.16 2690.79    -2.7 2705.79    1.06 2732.86    2.41
 2749.49    7.03 2758.21   10.92 2793.19      15 2803.18   17.18 2838.16   20.68
#Mann= 3 , 0 , 0
 1439.07    .055       0 1662.67   .0285       0 2758.21    .055       0
Bank Sta=1662.67,2758.21
XS Rating Curve= 0 ,0
Exp/Cntr(USF)=0.5,0.3
Exp/Cntr=0.3,0.1

Type RM Length L Ch R = 1 ,35173.12,734.97,1009.92,1301.42
XS GIS Cut Line= 2
360995.0328001215902233.47744978361462.0506267375900995.49208828
#Sta/Elev= 30
 1193.34   20.02 1208.32   10.47  1223.3   11.48 1238.28   17.37 1248.27   19.36
 1263.24   17.51 1273.23   17.69 1283.22   11.87  1293.2    8.75  1368.1    6.47
 1373.09    5.32 1393.06    8.05 1418.03    8.11 1433.01    5.91 1450.19    4.94
 1453.47    3.05 1473.72     .87 1550.69     .16 1581.39   -1.63 1869.74   -2.95
 2018.55   -1.47 2068.51   -2.94 2112.78     .47    2157    6.12 2186.96    11.3
 2271.85   15.31 2311.79   14.89 2336.76   18.41 2411.65   18.75 2516.51   24.15
#Mann= 3 , 0 , 0
 1193.34    .055       0 1418.03   .0285       0 2186.96    .055       0
Levee=-1,1274.11,17.58,-1,2339.14,18.55,,
Bank Sta=1418.03,2186.96
XS Rating Curve= 0 ,0
Exp/Cntr(USF)=0.5,0.3
Exp/Cntr=0.3,0.1

Type RM Length L Ch R = 1 ,34163.2 ,971.99,970.31,998.23
XS GIS Cut Line= 2
361840.6306077325902567.25777953362409.2559906375901643.65944352
#Sta/Elev= 30
 1239.56   26.48 1252.61   13.03 1267.31    3.21 1272.39    2.38  1283.1   -1.28
 1303.62   -4.72 1404.38   -2.47 1423.55   -3.08  1453.6   -1.25    1565    -.89
 1736.52     1.6    1740     4.8    1915     4.8 1920.35    1.14 2068.78   -3.97
  2071.5   -1.75 2077.66   -2.36 2079.42     .65 2091.27    -.83 2096.72    2.18
 2100.31     .86 2105.39    3.67 2114.25    3.04 2134.25    6.03 2164.23    7.31
 2229.21   14.05  2279.2   16.99 2304.19   16.96 2314.18   18.42 2324.18   21.42
#Mann= 5 ,-1 , 0
 1239.56    .055       0 1272.39   .0285       0    1740    .035       0
 1920.35   .0285       0 2105.39    .055       0
Bank Sta=1272.39,2105.39
XS Rating Curve= 0 ,0
Exp/Cntr(USF)=0.5,0.3
Exp/Cntr=0.3,0.1

Type RM Length L Ch R = 1 ,33192.89,1234.76,1006.17,727.63
XS GIS Cut Line= 2
362630.6979425485903133.15579225363408.9064251195901869.13893486
#Sta/Elev= 30
 1099.53   16.66 1193.52       2 1196.11     4.6 1246.29     4.6 1308.13   -3.16
  1349.2   -3.52 1390.19   -2.07 1575.04    -.56 1683.15    -3.5 1726.98    -.25
 1802.73    1.66 1812.54     4.6 1863.37     4.6 1872.25     .88 1884.47    1.69
 1895.18    4.45 1939.17    4.08 1954.16    6.24 2034.12    7.27  2079.1    6.59
 2096.62    2.79 2111.88    1.09 2201.93    -.08 2241.36    2.09 2264.03    5.45
 2363.98    6.08 2418.96   10.35 2503.92   13.76 2513.92   16.41 2583.89   20.76
#Mann= 4 ,-1 , 0
 1099.53    .024       0 1884.47    .035       0 2111.88   .0285       0
 2264.03    .055       0
Bank Sta=1099.53,2264.03
XS Rating Curve= 0 ,0
Exp/Cntr(USF)=0.5,0.3
Exp/Cntr=0.3,0.1

Type RM Length L Ch R = 1 ,32186.72,1219.67,994.54,671.77
XS GIS Cut Line= 2
 363631.709871595903578.71580343364207.1422299995902200.81437446
#Sta/Elev= 30
 1078.71   20.79 1083.71   17.56 1096.16    5.94 1101.62    2.87 1117.85    -.96
 1137.88   -3.17 1175.41   -1.49 1185.54    1.26 1396.22    1.17    1405     4.6
    1580     4.6 1591.57    1.65 1780.72    1.11  1840.6   -1.31 2044.77   -4.07
  2054.8     .27 2087.54    1.61 2197.18   -1.26 2222.78    2.19 2231.52    4.62
 2242.33    5.21 2302.25       8 2317.24   11.34  2347.2   13.93 2377.17   15.26
 2392.15   14.12  2432.1   17.17    2517   17.12 2541.97   19.97 2571.93   20.08
#Mann= 4 ,-1 , 0
 1078.71    .055       0    1405    .035       0 1591.57   .0285       0
 2242.33    .055       0
Bank Sta=1078.71,2242.33
XS Rating Curve= 0 ,0
Exp/Cntr(USF)=0.5,0.3
Exp/Cntr=0.3,0.1

Type RM Length L Ch R = 1 ,31192.18,1034.11,994.63,993.08
XS GIS Cut Line= 2
364659.094328575 5903964.7554875364993.4189005785902463.03305586
#Sta/Elev= 30
  624.39   24.61  634.38    12.2  645.88    2.99   649.4    2.03  674.61      .9
  735.88    1.37     740     4.5     950     4.5  955.84    1.47 1104.56     .61
 1199.53   -1.13 1209.85   -2.29  1259.6   -1.51 1285.02    2.02 1318.71    3.04
 1383.65    2.24    1390     4.5    1465     4.5 1466.49     .62 1748.66   -3.13
 1779.35   -2.75  1818.1    2.71 1822.53    4.68 1848.19    6.39 1873.17   10.08
 1953.09   13.56 1968.08   12.79 2008.04   14.86    2043   18.59 2162.88   21.46
#Mann= 6 ,-1 , 0
  624.39    .024       0     740    .035       0  955.84   .0285       0
 1285.02    .035       0 1466.49   .0285       0 1873.17    .055       0
Bank Sta=624.39,1873.17
XS Rating Curve= 0 ,0
Exp/Cntr(USF)=0.5,0.3
Exp/Cntr=0.3,0.1

Type RM Length L Ch R = 1 ,30197.55,1025.02,1021.21,1018.34
XS GIS Cut Line= 2
 365584.825019185904376.40324965366005.2681428385902487.85265764
#Sta/Elev= 30
  929.89   23.25  939.89   17.06 1074.88   10.78 1089.88   12.71 1139.87    9.05
 1154.87   10.07 1162.47     3.2 1186.24    -.28 1215.43   -1.19 1235.04     .36
 1248.87    -.87 1278.44    1.98 1398.24    2.02 1631.86   -1.52 1855.94    -.79
 2007.11    1.62    2012     4.2    2075     4.2 2079.76    1.67 2438.66    -.55
 2466.46    4.33 2514.71    3.83 2524.71    1.83 2554.71    3.72  2579.7    8.21
 2709.69    6.79 2724.69    4.04 2829.68   19.43 2849.67   18.71 2864.67   23.35
#Mann= 5 ,-1 , 0
  929.89    .055       0 1154.87   .0285       0    2012    .035       0
 2079.76   .0285       0  2579.7    .055       0
Levee=-1,920.97,25.37,-1,2611.08,8.23,,
Bank Sta=1154.87,2579.7
XS Rating Curve= 0 ,0
Exp/Cntr(USF)=0.5,0.3
Exp/Cntr=0.3,0.1

Type RM Length L Ch R = 1 ,29176.34,1138.34,976.42,790.73
XS GIS Cut Line= 2
366575.0504711595904614.59656991367048.7107041215902487.00490546
#Sta/Elev= 30
  874.87   20.36  889.87   13.16 1084.84   10.26 1114.84    6.38 1139.83    6.43
 1190.71    -.33 1215.73   -1.49 1343.76   -2.86 1433.44    1.35 1766.38      .2
 1944.53    1.49 1953.58    1.09    1960     4.3    2260     4.3 2268.33     .28
 2529.83   -1.24 2549.24     2.6 2559.62    9.31 2579.62   18.71 2614.62    16.3
  2694.6   16.48  2734.6    12.6 2784.59   11.93 2794.59    9.98 2839.58   10.46
 2874.58    8.06 2969.56    7.86 3004.56    8.69 3034.56   15.95 3054.55   25.68
#Mann= 5 ,-1 , 0
  874.87    .055       0 1139.83   .0285       0 1944.53    .035       0
 2268.33   .0285       0 2579.62    .055       0
Levee=-1,1080.27,10.49,-1,2581.21,18.28,,
Bank Sta=1139.83,2579.62
XS Rating Curve= 0 ,0
Exp/Cntr(USF)=0.5,0.3
Exp/Cntr=0.3,0.1

Type RM Length L Ch R = 1 ,28199.92,995.41,992.79,993.66
XS GIS Cut Line= 2
367655.3898128915904687.76428615367869.613936821  5902696.538264
#Sta/Elev= 30
   953.9    20.2  975.63     4.2  997.91   -1.82 1169.13    1.38 1179.25    -.27
 1246.03     .43 1256.19    1.76 1518.25    2.78 1563.64     .77 1675.29   -1.79
 1926.58    -.88 1946.78   -2.85 1956.78    -1.5 1966.78   -2.85 1977.19   -1.33
 2037.83    -.85 2078.12    1.05    2085     4.2    2229     4.2 2234.28     .63
 2527.66    -1.1 2556.52    1.83 2582.03   12.51 2646.95   11.34 2666.93    8.68
 2726.86    7.83 2891.66    8.75 2931.62   11.33  2946.6   16.44 2956.59   21.87
#Mann= 7 ,-1 , 0
   953.9    .055       0  975.63   .0285       0 1256.19    .035       0
 1563.64   .0285       0    2085    .035       0 2234.28   .0285       0
 2582.03    .055       0
Levee=0,,,-1,2598.63,12.92,,
Bank Sta=975.63,2582.03
XS Rating Curve= 0 ,0
Exp/Cntr(USF)=0.5,0.3
Exp/Cntr=0.3,0.1

Type RM Length L Ch R = 1 ,27207.13,1086.67,1005.59,915.85
XS GIS Cut Line= 2
 368658.787946125904640.07015667368841.4941561275902941.80450296
#Sta/Elev= 30
 1103.75   21.32 1139.49    3.95 1145.74    1.86    1150       4    1195       4
 1198.36    1.05 1408.78    -.79  1496.6    -.78 1575.28    1.33  1584.6    1.39
    1595       4    1900       4 1910.04    -.16 1937.86   -1.66 1999.01   -2.02
 2019.36   -3.44  2211.6    -.47 2462.69     .76  2483.4    2.51 2486.99    4.74
 2497.17    4.72 2512.16    2.32 2537.13     6.1  2567.1    6.52 2597.06    9.35
  2736.9   10.07 2751.89    10.8 2766.87   13.96 2796.84   16.56 2811.82   20.02
#Mann= 5 ,-1 , 0
 1103.75    .055       0 1139.49   .0285       0 1575.28    .035       0
 1910.04   .0285       0 2486.99    .055       0
Bank Sta=1139.49,2486.99
XS Rating Curve= 0 ,0
Exp/Cntr(USF)=0.5,0.3
Exp/Cntr=0.3,0.1

Type RM Length L Ch R = 1 ,26201.55,1068.28,1001.65,945.48
XS GIS Cut Line= 2
369693.6218208885904800.33809111369798.5638235755902765.25934895
#Sta/Elev= 30
 1053.86   20.02 1073.83    7.09 1078.83    5.54 1143.76    4.96    1310     .94
    1315     3.9    1645     3.9 1648.78     1.8 1662.12    1.19 1805.22    1.25
 2007.26   -2.55 2128.61    -.65 2271.01    -.94  2382.8   -4.74 2421.41    2.21
 2432.36    9.08 2537.25   11.55  2677.1   10.36 2687.08     7.4 2727.04    1.43
    2767    2.03 2811.95    9.45  2856.9    7.93 2876.88    2.99 2971.78    3.56
 2991.76    4.38 3011.74    7.77 3056.69    9.52 3081.66    15.1 3091.65   20.19
#Mann= 5 ,-1 , 0
 1053.86    .055       0 1143.76   .0285       0    1315    .035       0
 1662.12   .0285       0 2432.36    .055       0
Levee=0,,,-1,2548.85,11.54,,
Bank Sta=1143.76,2432.36
XS Rating Curve= 0 ,0
Exp/Cntr(USF)=0.5,0.3
Exp/Cntr=0.3,0.1

Type RM Length L Ch R = 1 ,25199.9 ,1065.31,998.49,975.09
XS GIS Cut Line= 2
370718.7755874455905151.77759483370740.4105410685903303.20609274
#Sta/Elev= 30
  804.43   24.63  829.41    8.17   839.4    5.94 1184.16       5 1229.12    3.88
 1274.09     5.7 1314.06    4.15 1329.05    4.57 1349.04    8.34 1360.51    5.88
 1388.08   -3.66 1437.24    -.43 1498.09     .38 1517.74   -1.69 1558.29   -1.98
 1708.49    1.11 1991.75    1.07 2032.18     .62 2052.44   -2.87 2072.87   -4.74
 2185.69   -1.71 2443.79   -2.34 2454.04   -1.42 2472.27    2.81 2498.22    6.52
 2508.21    5.64  2528.2    6.77 2553.18   10.38 2583.16   11.19 2653.11   20.85
#Mann= 5 ,-1 , 0
  804.43    .055       0 1349.04   .0285       0 1708.49   .0285       0
 1991.75   .0285       0 2498.22    .055       0
Levee=-1,1347.83,9.11,0,,,,
#XS Ineff= 2 , 0
       0  1016.5      11               0
Permanent Ineff=
       F       F
Bank Sta=1349.04,2498.22
XS Rating Curve= 0 ,0
Exp/Cntr(USF)=0.5,0.3
Exp/Cntr=0.3,0.1

Type RM Length L Ch R = 1 ,24201.41,139.37,137.37,138.3
XS GIS Cut Line= 2
371755.4124039625905315.34396905371721.1203393415903600.74243302
#Sta/Elev= 30
  779.98   21.17  809.97    6.19  819.97    4.88 1324.96    4.42 1339.96    6.06
 1444.95    5.35 1454.95    8.87 1549.95   10.06 1559.95    6.52 1653.94    -2.6
  1787.9    -2.2  1797.9   -4.02  1858.7   -2.02 1956.68   -5.99 2017.59   -5.53
 2037.37  -13.16 2066.03  -20.38 2096.55  -18.89 2126.27   -8.67 2136.02   -7.56
 2155.63  -14.19 2185.55  -14.09 2204.82   -11.1 2224.98  -12.08 2265.34   -5.53
 2363.69   -2.14 2405.55    3.26 2429.92    3.24 2454.92   15.56 2494.92   20.43
#Mann= 3 , 0 , 0
  779.98    .055       0 1549.95   .0285       0 2454.92    .055       0
Levee=-1,1535.47,9.67,-1,2478.53,18.01,,
#XS Ineff= 2 , 0
       0    2015      11    2375       0      11
Permanent Ineff=
       F       F
Bank Sta=1549.95,2454.92
XS Rating Curve= 0 ,0
Exp/Cntr(USF)=0.5,0.3
Exp/Cntr=0.3,0.1
